HEC-RAS study GeorgesCreek.prj: Georges Creek Limited Detail Study

--- GeorgesCreek.g06 (geometry) --- (continued)

Type RM Length L Ch R = 1 ,49497   ,437,437,437
BEGIN DESCRIPTION:
Georges Creek 99.0
END DESCRIPTION:
XS GIS Cut Line= 3
      1522126.63      1100204.38      1522147.74      1099656.99
      1522046.25      1099428.72
#Sta/Elev= 22
  4618.3  952.26  4628.3  950.88  4660.8  947.21  4740.8   936.7  4743.3  936.47
  4766.5  928.13    4780  930.75  4783.3  931.54    4789  932.61  4803.3   932.4
  4875.4  928.06  4943.7  932.39  4968.8  934.93  4994.5  928.06  4995.5  926.06
  5004.5  926.06  5005.5  928.06  5025.5  935.46  5125.1  934.72  5163.8  941.74
  5210.4  951.35  5236.9  955.07
#Mann= 3 ,-1,0
  4618.3     .14       0  4994.5     .05       0  5005.5     .15       0
Bank Sta=4994.5,5005.5
XS Rating Curve= 0 ,0
Exp/Cntr=0.3,0.1

Type RM Length L Ch R = 1 ,49060   ,563,563,563
BEGIN DESCRIPTION:
Georges Creek 98.0
END DESCRIPTION:
XS GIS Cut Line= 3
      1522383.84      1100204.38      1522600.86      1099629.67
      1522749.57       1099444.8
#Sta/Elev= 19
  4803.5  952.02  4860.9  945.36  4865.5  944.54  4909.6  932.24  4924.2  929.18
  4927.5  927.86  4949.8  933.55  4974.6  933.65  4994.5  927.86  4995.5  925.86
  5004.5  925.86  5005.5  927.86  5006.5  929.91  5020.2  933.55  5072.9  931.78
  5113.8  930.06  5265.4  949.41  5279.5  952.19  5284.3  952.76
#Mann= 3 ,-1,0
  4803.5     .15       0  4994.5     .05       0  5005.5     .15       0
Bank Sta=4994.5,5005.5
XS Rating Curve= 0 ,0
Exp/Cntr=0.3,0.1

Type RM Length L Ch R = 1 ,48497   ,473,473,473
BEGIN DESCRIPTION:
Georges Creek 97.0
END DESCRIPTION:
XS GIS Cut Line= 3
      1523589.53      1099959.23      1522988.77      1099563.69
        1522825.        1099425.
#Sta/Elev= 27
    4297  962.29  4338.5  938.58  4341.4  937.58    4398  931.12  4398.9  931.07
  4714.5  930.54  4884.1  928.95  4887.5  929.26  4904.9  929.52  4922.7  932.11
  4954.2  935.99  4965.1  936.99    4967  937.16  4982.9  932.43  4992.1  929.42
    4994     927  4995.1     925    5005     925  5006.1     927  5036.7  943.86
  5131.6  947.71  5139.4  948.46  5147.1  949.78  5152.5  950.53  5160.7  948.52
  5213.8  963.11  5214.6  963.23
#Mann= 4 ,-1,0
    4297      10       0  4965.1     .15       0    4994     .05       0
  5006.1     .15       0
Bank Sta=4994,5006.1
XS Rating Curve= 0 ,0
Exp/Cntr=0.5,0.3

Type RM Length L Ch R = 1 ,48024   ,102,102,102
BEGIN DESCRIPTION:
Georges Creek 96.0
END DESCRIPTION:
XS GIS Cut Line= 3
      1523702.06      1099693.97      1523320.26      1099199.64
      1522994.72       1099042.9
#Sta/Elev= 25
  4294.5  944.27  4311.6  938.66  4350.2   929.7  4523.4  928.45  4545.3  928.99
  4623.8  929.19  4625.8  929.26  4731.5  932.01  4736.3  932.04  4820.8  935.75
  4879.1  934.31  4890.9  934.77  4906.2  935.01  4919.8  934.41  4943.3  935.62
  4961.8  936.04    4985  931.76    4991  925.76    5009  925.76    5015  931.76
    5024  933.39  5147.4  951.43  5173.8  954.18  5179.4  954.63  5186.3  953.99
#Mann= 3 ,-1,0
  4294.5     .14       0    4985    .049       0    5015     .14       0
#XS Ineff= 2 , 0
            4931     943    5069          947.08
Permanent Ineff=
       F       F
Bank Sta=4985,5015
XS Rating Curve= 0 ,0
Exp/Cntr=0.5,0.3

Type RM Length L Ch R = 3 ,47970   ,,,
BEGIN DESCRIPTION:
Jordan Rd. (Georges Cr.) - TOR
Structure ID: Jordan Rd. (Georges Cr.)
Approximate Survey Structure
END DESCRIPTION:
Bridge Culvert--1,0,-1,-1, 0
Deck Dist Width WeirC Skew NumUp NumDn MinLoCord MaxHiCord MaxSubmerge Is_Ogee
39,30,3,0, 24, 24, , , , 0, 1,1,,
  4244.5  4261.3  4274.8  4277.2    4285    4970    4970    5030    5030  5039.2
  5041.5  5047.8  5050.5    5052  5064.9  5072.8  5078.2  5140.1  5140.5  5181.9
  5183.5  5194.2  5210.4  5259.1
  955.54  951.09  947.12  945.53     943     943     943     943     943     943
  943.24  943.19   944.6   944.9  946.63   947.5     947  949.88  949.87  954.18
  954.31  953.33  956.87  961.66
  905.76  905.76  905.76  905.76  905.76  905.76     942     942  905.76  905.76
  905.76  905.76  905.76  905.76  905.76  905.76  905.76  905.76  905.76  905.76
  905.76  905.76  905.76  905.76
  4244.5  4261.3  4274.8  4277.2    4285    4970    4970    5030    5030  5039.2
  5041.5  5047.8  5050.5    5052  5064.9  5072.8  5078.2  5140.1  5140.5  5181.9
  5183.5  5194.2  5210.4  5259.1
  955.54  951.09  947.12  945.53     943     943     943     943     943     943
  943.24  943.19   944.6   944.9  946.63   947.5     947  949.88  949.87  954.18
  954.31  953.33  956.87  961.66
  905.76  905.76  905.76  905.76  905.76  905.76     942     942  905.76  905.76
  905.76  905.76  905.76  905.76  905.76  905.76  905.76  905.76  905.76  905.76
  905.76  905.76  905.76  905.76
Pier Skew, UpSta & Num, DnSta & Num=  ,4985, 2 ,4985, 2 , 0 , 0 , 0 ,0,0
       1       1
     938     942
       1       1
  937.75     942
Pier Skew, UpSta & Num, DnSta & Num=  ,5015, 2 ,5015, 2 , 0 , 0 , 0 ,0,0
       1       1
     938     942
       1       1
  937.75     942
Abutment Skew #Up #Dn= , 2 , 2
    4970  4972.5
     942  936.94
    4970  4972.5
     942  931.59
Abutment Skew #Up #Dn= , 2 , 2
  5027.5    5030
  934.85     942
  5027.5    5030
  934.04     942
BR Coef=-1 ,-1 , 0 ,1.25, 0 ,,,0.8,0,2,0,
WSPro=,,,, 1 ,,,, 0 ,,,, 0 ,,,,-1 ,-1 ,-1 , 0 , 0 , 0 , 0 , 0
BC Design=,, 0 ,, 0 ,,,,,,
BC HTab HWMax=954.63
BC Use User HTab Curves=0
BC User HTab FreeFlow(D)= 0

Type RM Length L Ch R = 1 ,47922   ,492,492,492
BEGIN DESCRIPTION:
Georges Creek 95.5
END DESCRIPTION:
XS GIS Cut Line= 3
      1523754.31      1099633.69      1523396.62      1099111.22
      1523034.91      1098974.58
#Sta/Elev= 30
  4232.6  946.54  4261.9  938.48  4290.2   931.6  4295.7   929.7  4315.4  927.86
    4333  927.35  4421.6  928.35  4479.9  927.09  4535.3  930.16  4617.6  928.72
  4660.2  929.91    4673  931.48  4688.6   932.1  4723.6  932.29    4735  931.94
  4782.9  935.02  4888.5  935.84    4914  936.55  4925.5   934.5  4946.2  934.39
    4985  930.51    4991  925.51    5009  925.51    5015  930.51  5022.1  931.71
    5042  940.29  5075.4  944.38  5094.2  946.01  5192.7   952.8  5252.5   959.3
#Mann= 3 ,-1,0
  4232.6     .14       0    4985    .049       0    5015     .14       0
#XS Ineff= 2 , 0
            4937     943    5063          946.38
Permanent Ineff=
       F       F
Bank Sta=4985,5015
XS Rating Curve= 0 ,0
Exp/Cntr=0.5,0.3

Type RM Length L Ch R = 1 ,47430   ,427,427,427
BEGIN DESCRIPTION:
Georges Creek 95.0
END DESCRIPTION:
XS GIS Cut Line= 3
       1523794.5      1099673.88       1523688.6      1098941.61
      1523975.59      1098606.78
#Sta/Elev= 30
  4255.7  956.36  4342.9   929.7    4424  926.82  4438.5  926.75  4450.2  927.84
  4498.6  929.59  4556.4  925.79  4613.3  929.23  4736.3  925.98  4746.9  926.24
  4761.8  928.43  4775.1  926.99  4794.5  925.89    4847  927.62  4871.4  927.67
  4903.8  926.14    4924  926.18    4963  927.04  4983.7  925.67    4994  924.11
  4995.1  922.11    5005  922.11  5006.1  924.11  5067.6  927.55  5130.9  933.05
    5202  941.31  5206.8  941.47  5245.6  945.36  5288.4  946.99  5320.9     954
#Mann= 3 ,-1,0
  4255.7     .14       0    4994    .049       0  5006.1     .14       0
Bank Sta=4994,5006.1
XS Rating Curve= 0 ,0
Exp/Cntr=0.3,0.1

Type RM Length L Ch R = 1 ,47003   ,553,553,553
BEGIN DESCRIPTION:
Georges Creek 94.0
END DESCRIPTION:
XS GIS Cut Line= 3
       1523923.1      1099685.94      1524002.17      1099239.24
      1524204.13       1098936.3
#Sta/Elev= 17
  4495.4  951.21  4572.3  932.73  4663.9   929.7  4853.4  928.33  4915.6  929.51
    4949  929.93  4959.1  929.65  4994.5  924.11  4995.5  922.11  5004.5  922.11
  5005.5  924.11  5006.6  924.11  5048.7  929.26  5118.2  932.81    5146  931.26
  5168.4  937.66  5214.6  953.35
#Mann= 3 ,-1,0
  4495.4     .14       0  4994.5    .049       0  5005.5     .14       0
Bank Sta=4994.5,5005.5
XS Rating Curve= 0 ,0
Exp/Cntr=0.3,0.1

Type RM Length L Ch R = 1 ,46450   ,453,453,453
BEGIN DESCRIPTION:
Georges Creek 93.0
END DESCRIPTION:
XS GIS Cut Line= 3
      1524352.95      1099797.29      1524496.44      1099494.35
      1524570.85      1099058.54
#Sta/Elev= 29
  4767.8  949.46  4829.6  939.18  4869.6  931.32  4873.7  930.66  4905.8  926.71
  4969.8   920.9  4974.1  920.48  4990.9  920.35    4994  920.26  4995.1  918.26
    5005  918.26  5006.1  920.26  5036.2  921.28  5042.8  921.61  5054.6  921.28
  5055.2  921.29  5125.1  920.39  5132.1  920.49  5134.6  920.45  5173.6  921.49
  5183.3  923.53  5201.3  925.67  5232.6  928.05  5265.3  933.06  5284.5  933.81
  5292.4  937.02  5355.2  949.35  5358.7  949.79  5360.7  950.29
#Mann= 3 ,-1,0
  4767.8     .14       0    4994    .049       0  5006.1     .14       0
Bank Sta=4994,5006.1
XS Rating Curve= 0 ,0
Exp/Cntr=0.3,0.1

Type RM Length L Ch R = 1 ,45997   ,674,674,674
BEGIN DESCRIPTION:
Georges Creek 92.0
END DESCRIPTION:
XS GIS Cut Line= 3
      1524703.72      1100068.35      1524910.97      1099621.88
      1525267.09      1099276.44
#Sta/Elev= 28
  4628.3  946.09  4668.6  942.53  4683.2   942.2  4747.8  932.98  4751.3  932.82
  4757.3  932.01  4759.9  931.74  4833.8  922.63  4918.3  917.54  4964.2  916.68
  4977.4   917.6    4994  915.82  4995.1  913.82    5005  913.82  5006.1  915.82
  5113.2  920.98  5213.3  915.85  5214.2  915.82  5216.7  915.87  5217.2  915.93
  5218.6     916  5218.8  916.13  5219.5  916.24  5273.8  921.84  5283.2   922.1
  5348.8  929.97  5398.2  939.05  5427.6  943.66
#Mann= 3 ,-1,0
  4628.3    .125       0    4994    .048       0  5006.1     .15       0
Bank Sta=4994,5006.1
XS Rating Curve= 0 ,0
Exp/Cntr=0.3,0.1

Type RM Length L Ch R = 1 ,45323   ,862,862,862
BEGIN DESCRIPTION:
Georges Creek 91.0
END DESCRIPTION:
XS GIS Cut Line= 3
        1525198.      1100148.07      1525463.74      1099972.68
       1525559.4      1099499.66
#Sta/Elev= 30
  4787.9     940  4797.3  939.03  4824.5  934.81  4843.3   933.6  4870.1  931.26
  4890.1   930.4  4899.8  929.67  4923.1  926.51  4946.1  922.81  4954.6  922.13
  4958.1  921.76  4970.6  920.18    4994  912.64  4995.1  910.64    5005  910.64
  5006.1  912.64  5015.7  916.08  5024.1  917.79  5081.8  919.11  5172.8  917.85
  5238.2  926.05  5260.3  926.47  5273.1  926.26  5298.4  929.33  5302.4  930.28
  5308.3  931.34  5376.5  940.07  5393.8  937.08  5402.9  943.66  5407.3  944.51
#Mann= 3 ,-1,0
  4787.9    .125       0    4994    .048       0  5006.1     .15       0
Bank Sta=4994,5006.1
XS Rating Curve= 0 ,0
Exp/Cntr=0.3,0.1

Type RM Length L Ch R = 1 ,44461   ,464,464,464
BEGIN DESCRIPTION:
Georges Creek 89.0
END DESCRIPTION:
XS GIS Cut Line= 3
      1525506.26      1100631.72      1525857.03        1100265.
      1526165.29      1100243.74
#Sta/Elev= 30
  4378.1  926.48  4407.9  924.57  4420.6  922.88  4428.8     923  4434.9  922.61
  4533.3  919.25  4543.7  919.24  4572.2   918.4  4585.7  918.51    4620  914.37
  4651.3  914.34  4658.1   914.5  4671.6   914.1    4707  914.62  4709.7  914.17
  4725.8  910.64    4735   913.2  4743.8  915.87    4783  915.37  4880.5  914.11
  4977.4  915.03    4994  910.08  4995.1  908.08    5005  908.08  5006.1  910.08
  5018.5  916.39    5031  920.97  5083.1  936.08  5094.2  939.99  5102.3  941.36
#Mann= 4 ,-1,0
  4378.1      10       0    4783    .125       0    4994    .048       0
  5006.1     .15       0
Bank Sta=4994,5006.1
XS Rating Curve= 0 ,0
Exp/Cntr=0.3,0.1

Type RM Length L Ch R = 1 ,43997   ,500,500,500
BEGIN DESCRIPTION:
Georges Creek 88.0
END DESCRIPTION:
XS GIS Cut Line= 3
        1525625.        1101025.      1526161.23      1100669.69
      1526340.68      1100583.88
#Sta/Elev= 26
  4356.7     935  4375.8  933.61  4402.9  931.02  4432.6  926.95  4466.3  924.63
  4502.9  919.64  4506.5  919.26  4530.4  917.29  4565.2  917.39  4587.6  914.01
  4637.6  912.01  4639.6     912  4640.8  911.73  4653.3   909.4  4666.8  911.68
  4674.9  913.35  4675.1  913.34    4693  912.66  4993.4  909.12  4994.6  907.12
  5005.4  907.12  5006.6  909.12  5017.7  909.12  5042.8     918  5091.9  929.41
  5140.1  939.43
#Mann= 4 ,-1,0
  4356.7      10       0  4675.1    .125       0  4993.4    .048       0
  5006.6     .15       0
Bank Sta=4993.4,5006.6
XS Rating Curve= 0 ,0
Exp/Cntr=0.3,0.1

Type RM Length L Ch R = 1 ,43497   ,500,500,500
BEGIN DESCRIPTION:
Georges Creek 87.0
END DESCRIPTION:
XS GIS Cut Line= 3
      1526457.61       1101630.9      1526494.17      1101030.89
        1526625.        1100825.
#Sta/Elev= 28
  4398.9     944    4467  932.65  4467.8  932.58  4545.6  924.86  4620.1  919.01
  4639.3  915.28  4645.4  913.83  4651.3  915.81  4658.1  918.39  4714.8  911.43
    4800  909.41    4823  908.86  4851.6  904.44  4854.5  905.66  4869.6  911.77
  4903.2     911  4961.7  911.21  4977.1  911.58  4992.9  904.44  4993.9  902.44
  5006.1  902.44  5007.1  904.44  5010.9  908.21  5040.2  914.37  5101.5  924.81
  5121.1  927.47  5151.7  934.87  5221.8  948.33
#Mann= 4 ,-1,0
  4398.9      10       0    4800    .125       0  4992.9    .048       0
  5007.1     .15       0
Bank Sta=4992.9,5007.1
XS Rating Curve= 0 ,0
Exp/Cntr=0.3,0.1

Type RM Length L Ch R = 1 ,42997   ,543,543,543
BEGIN DESCRIPTION:
Georges Creek 86.0
END DESCRIPTION:
XS GIS Cut Line= 3
        1527025.        1101625.       1526980.1      1101070.45
      1526909.36      1100865.57
#Sta/Elev= 29
  4443.6  934.53    4477  928.67  4522.1  922.89  4597.5  914.66  4607.5  912.44
  4609.8   911.4  4610.9  911.69    4623  916.37  4639.6  914.48  4646.6  913.19
  4725.3  906.28  4728.3  906.15  4751.5  902.87  4767.1  908.55  4841.9  911.29
  4963.2  909.57  4974.8  909.71  4983.8  908.17  4992.9  904.06  4993.9  902.06
  5006.1  902.06  5007.1  904.06  5023.6  910.33  5034.8  913.58  5047.2   916.7
  5054.8  917.77  5084.8  923.36    5111  926.04  5216.8  941.83
#Mann= 4 ,-1,0
  4443.6      10       0  4841.9    .125       0  4992.9    .048       0
  5007.1     .15       0
Bank Sta=4992.9,5007.1
XS Rating Curve= 0 ,0
Exp/Cntr=0.3,0.1

Type RM Length L Ch R = 1 ,42454   ,457,457,457
BEGIN DESCRIPTION:
Georges Creek 85.0
END DESCRIPTION:
XS GIS Cut Line= 3
      1527371.75      1101609.64      1527419.58      1101248.23
       1527605.6       1101019.7
#Sta/Elev= 29
  4557.5  926.94  4568.3  924.84  4652.6  915.37    4656   913.3    4665  908.36
  4673.2  910.25  4673.7  910.35  4676.3  910.88  4686.6  909.44  4715.7  905.78
  4719.4  904.73  4724.4  903.93  4731.5  904.38  4737.2  904.91  4743.4  906.26
    4800  906.37    4801  906.37  4801.5  906.36  4907.8  906.63    4910  906.75
  4922.1  906.96  4971.7  907.96  4976.6  907.17  4992.9  903.64  4993.9  901.64
  5006.1  901.64  5007.1  903.64  5020.1  910.44  5167.4  939.76
#Mann= 4 ,-1,0
  4557.5      10       0    4800    .125       0  4992.9    .048       0
  5007.1     .15       0
Bank Sta=4992.9,5007.1
XS Rating Curve= 0 ,0
Exp/Cntr=0.3,0.1

Type RM Length L Ch R = 1 ,41997   ,500,500,500
BEGIN DESCRIPTION:
Georges Creek 84.0
END DESCRIPTION:
XS GIS Cut Line= 3
       1527605.6      1101726.56      1527875.94      1101344.76
      1527866.03      1101184.46
#Sta/Elev= 19
    4588   927.8  4603.4  925.65    4672   913.9  4684.2  908.61  4703.6  907.86
  4747.8  903.97  4771.1  900.23    4792  905.49    4800  905.24    4838  904.03
    4929  906.37  4980.1  905.89  4992.9  900.23  4993.9  898.23  5006.1  898.23
  5007.1  900.23  5027.6  908.09  5097.8  926.67  5105.1  928.39
#Mann= 4 ,-1,0
    4588      10       0    4800    .125       0  4992.9    .048       0
  5007.1     .15       0
Bank Sta=4992.9,5007.1
XS Rating Curve= 0 ,0
Exp/Cntr=0.3,0.1

Type RM Length L Ch R = 1 ,41497   ,500,500,500
BEGIN DESCRIPTION:
Georges Creek 83.0
END DESCRIPTION:
XS GIS Cut Line= 3
       1528360.3      1102236.79      1528364.69      1101408.04
        1528425.        1101225.
#Sta/Elev= 28
  4219.3  927.33  4226.5  925.78  4233.1  923.79    4306   905.8  4320.6  906.11
  4396.1  905.53  4397.8  905.45  4420.2  902.49  4434.9  904.81  4443.6  904.62
    4480  905.02  4482.2  905.04  4663.8  900.23  4726.4  902.15  4731.4  901.22
    4745  896.97  4749.3  898.45    4757  900.74  4761.6  902.39  4808.7  901.38
  4868.7  902.07  4929.1  904.32    4980  904.04  4992.9  896.97  4993.9  894.97
  5006.1  894.97  5007.1  896.97  5139.2  924.74
#Mann= 4 ,-1,0
  4219.3      10       0    4480    .125       0  4992.9    .048       0
  5007.1     .15       0
Bank Sta=4992.9,5007.1
XS Rating Curve= 0 ,0
Exp/Cntr=0.3,0.1

Type RM Length L Ch R = 1 ,40997   ,593,593,593
BEGIN DESCRIPTION:
Georges Creek 82.0
END DESCRIPTION:
XS GIS Cut Line= 3
      1528727.02      1102188.95      1528803.81      1101205.24
      1528796.12      1101030.33
#Sta/Elev= 30
  4013.3  928.32  4035.9  927.68  4098.1   924.6  4119.9  922.75  4152.9   922.6
  4177.5  919.89  4200.1  915.24  4236.2  908.91  4270.2   900.6    4284  896.38
  4289.1  897.45  4293.9  897.18  4296.9  897.75  4301.8  897.92  4327.2  896.95
  4331.3  896.51  4352.6  901.41  4442.2  900.83    4600  902.91  4749.8  898.79
  4880.1  901.94  4930.5  901.88  4967.9  902.51  4984.7  902.21  4992.9  896.38
  4993.9  894.38  5006.1  894.38  5007.1  896.38  5056.8  909.56  5118.2  926.73
#Mann= 4 ,-1,0
  4013.3      10       0    4600    .125       0  4992.9    .048       0
  5007.1     .15       0
Bank Sta=4992.9,5007.1
XS Rating Curve= 0 ,0
Exp/Cntr=0.3,0.1

Type RM Length L Ch R = 1 ,40404   ,407,407,407
BEGIN DESCRIPTION:
Georges Creek 81.0
END DESCRIPTION:
XS GIS Cut Line= 4
      1529205.36      1102130.49      1529290.39      1101375.79
      1529449.84      1101211.03      1529625.22      1101115.36
#Sta/Elev= 30
  4113.1  923.26  4120.4   922.8  4134.9  922.55  4164.6  920.63  4174.9  920.13
  4205.7  916.11  4235.7  914.09  4334.4  900.81  4341.3  900.71  4426.6  894.68
  4436.2  896.54  4449.1  899.49    4600  898.93    4848  898.02  4872.6  898.47
  4972.1   899.3  4976.1  899.06  4981.8  897.86  4992.2   894.4  4993.3   892.4
  5006.7   892.4  5007.8   894.4    5010   895.7  5017.7  896.21  5031.7  900.37
    5061  906.36  5101.9   911.7  5126.7  915.37  5145.1  916.77  5162.5  918.22
#Mann= 4 ,-1,0
  4113.1      10       0    4600    .125       0  4992.2    .048       0
  5007.8     .15       0
Bank Sta=4992.2,5007.8
XS Rating Curve= 0 ,0
Exp/Cntr=0.3,0.1

Type RM Length L Ch R = 1 ,39997   ,500,500,500
BEGIN DESCRIPTION:
Georges Creek 80.0
END DESCRIPTION:
XS GIS Cut Line= 3
        1529425.        1102225.      1529607.37      1101594.32
        1529825.        1101425.
#Sta/Elev= 27
  4343.5  927.95  4372.6  923.39    4391  921.03  4395.2  920.32  4470.2  900.78
  4485.8  899.11  4548.4  895.59  4603.2  896.06  4628.5  896.86  4656.2  892.84
  4671.2  897.75  4757.7   899.2  4758.8  899.22  4781.6  899.07  4890.4     896
  4992.1   896.3  4992.9  892.84  4993.9  890.84  5006.1  890.84  5007.1  892.84
  5014.9  893.56  5042.6  898.97  5061.6  900.82    5085  903.75  5093.5  905.14
  5107.8  908.39  5156.5  922.84
#Mann= 4 ,-1,0
  4343.5      10       0  4757.7    .125       0  4992.9    .048       0
  5007.1     .15       0
Bank Sta=4992.9,5007.1
XS Rating Curve= 0 ,0
Exp/Cntr=0.3,0.1

Type RM Length L Ch R = 1 ,39497   ,812,812,812
BEGIN DESCRIPTION:
Georges Creek 79.0
END DESCRIPTION:
XS GIS Cut Line= 3
      1529868.38      1102335.11      1529979.96      1101915.66
      1530099.57      1101715.94
#Sta/Elev= 24
    4566  940.05  4567.3   939.6  4695.3  906.99  4724.6  903.27    4763  899.96
  4784.6  896.94  4792.5  894.64  4804.3  891.57  4837.7  894.63  4946.1  894.89
  4980.9  894.29  4992.9  891.29  4993.9  889.29  5006.1  889.29  5007.1  891.29
  5021.9  901.85    5059  899.44    5093  908.26  5104.4  911.49  5130.7  922.22
    5146  924.41  5153.1     925  5225.6  940.42  5232.8  940.69
#Mann= 3 ,-1,0
    4566    .125       0  4992.9    .048       0  5007.1     .15       0
Bank Sta=4992.9,5007.1
XS Rating Curve= 0 ,0
Exp/Cntr=0.5,0.3

Type RM Length L Ch R = 1 ,38685   ,155,155,155
BEGIN DESCRIPTION:
Georges Creek 78.0
END DESCRIPTION:
XS GIS Cut Line= 4
       1530702.8      1102712.46      1530639.02      1102374.97
      1530623.08      1102157.06       1530665.6      1101859.43
#Sta/Elev= 30
  4610.9  927.17  4672.8  920.25  4691.5  916.49  4710.5  914.15    4725  910.99
    4742  910.72  4766.6  908.57  4794.7     908  4841.5  901.52  4883.1  899.24
  4965.6  897.25  4980.8     895  4990.4   885.2  5009.7   885.2  5019.3     895
  5077.7     895  5084.3   894.5  5131.6  895.56  5172.8  894.14  5211.9  894.17
  5233.4  893.16    5287  894.85  5299.8  895.98  5315.1   895.8  5343.1  898.91
  5365.3  899.61  5414.4  896.83  5419.3  897.64  5438.9  904.31  5457.1   908.5
#Mann= 3 ,-1,0
  4610.9     .15       0  4980.8    .048       0  5019.3    .135       0
#XS Ineff= 2 , 0
          4920.5  902.76  5079.5          900.92
Permanent Ineff=
       F       F
Bank Sta=4980.8,5019.3
XS Rating Curve= 0 ,0
Exp/Cntr=0.5,0.3

Type RM Length L Ch R = 3 ,38628   ,,,
BEGIN DESCRIPTION:
Grant Valley Rd. - TOR
Structure ID: LDS_GC_11
Approximate Survey Structure
END DESCRIPTION:
Bridge Culvert--1,0,-1,-1, 0
Deck Dist Width WeirC Skew NumUp NumDn MinLoCord MaxHiCord MaxSubmerge Is_Ogee
39.5,35,3,0, 20, 20, , , , 0, 1,1,,
  4647.7  4765.5  4882.4    4960    4960    5040    5040  5137.6  5138.4    5149
  5159.2    5192  5228.4  5334.1  5390.9  5397.1  5401.3  5417.9  5435.8  5437.3
   915.7  907.49  904.46     901     901     901     901  900.79   900.8  900.72
  900.89  900.56  900.62  903.52  906.24  906.18     906  909.15  908.95  909.07
   865.2   865.2   865.2   865.2   899.5   899.5   865.2   865.2   865.2   865.2
   865.2   865.2   865.2   865.2   865.2   865.2   865.2   865.2   865.2   865.2
  4647.7  4765.5  4882.4    4960    4960    5040    5040  5137.6  5138.4    5149
  5159.2    5192  5228.4  5334.1  5390.9  5397.1  5401.3  5417.9  5435.8  5437.3
   915.7  907.49  904.46     901     901     901     901  900.79   900.8  900.72
  900.89  900.56  900.62  903.52  906.24  906.18     906  909.15  908.95  909.07
   865.2   865.2   865.2   865.2   899.5   899.5   865.2   865.2   865.2   865.2
   865.2   865.2   865.2   865.2   865.2   865.2   865.2   865.2   865.2   865.2
Pier Skew, UpSta & Num, DnSta & Num=  ,4980, 2 ,4980, 2 , 0 , 0 , 0 ,0,0
       1       1
  894.37   899.5
       1       1
  889.84   899.5
Pier Skew, UpSta & Num, DnSta & Num=  ,5020, 2 ,5020, 2 , 0 , 0 , 0 ,0,0
       1       1
  896.14   899.5
       1       1
  895.68   899.5
Abutment Skew #Up #Dn= , 2 , 2
    4960    4963
   899.5  897.28
    4960    4963
   899.5  892.74
Abutment Skew #Up #Dn= , 2 , 2
    5037    5040
  895.08   899.5
    5037    5040
  895.04   899.5
BR Coef=-1 ,-1 , 0 ,1.25, 0 ,,,0.8,0,2,0,
WSPro=,,,, 1 ,,,, 0 ,,,, 0 ,,,,-1 ,-1 ,-1 , 0 , 0 , 0 , 0 , 0
BC Design=,, 0 ,, 0 ,,,,,,
BC HTab HWMax=927.17
BC Use User HTab Curves=0
BC User HTab FreeFlow(D)= 0

Type RM Length L Ch R = 1 ,38530   ,533,533,533
BEGIN DESCRIPTION:
Georges Creek 77.0
END DESCRIPTION:
XS GIS Cut Line= 3
      1530851.61      1102720.43      1530769.23      1102268.67
      1530833.01      1101907.27
#Sta/Elev= 27
  4633.7  913.24  4685.6  907.82  4747.3   902.9  4785.6  896.01  4797.8  896.07
  4820.9  894.81  4856.7  894.27  4896.3     890  4898.1  890.19  4901.5  890.36
  4904.8   890.4  4912.7  890.07  4951.7  893.57  4954.3  893.72  4964.7  892.55
  4980.8  893.05  4990.4  884.95  5009.7  884.95  5019.3  893.05  5092.9  894.41
  5144.4  892.97  5285.6  896.06  5330.3  900.02    5413  912.86  5426.7  914.54
  5452.4  919.06  5459.9  920.02
#Mann= 3 ,-1,0
  4633.7     .15       0  4980.8    .048       0  5019.3    .135       0
#XS Ineff= 2 , 0
          4879.5  904.54  5120.5          900.83
Permanent Ineff=
       F       F
Bank Sta=4980.8,5019.3
XS Rating Curve= 0 ,0
Exp/Cntr=0.5,0.3

Type RM Length L Ch R = 1 ,37997   ,500,500,500
BEGIN DESCRIPTION:
Georges Creek 76.0
END DESCRIPTION:
XS GIS Cut Line= 3
        1531225.        1102825.      1531289.22      1102515.03
        1531425.        1102025.
#Sta/Elev= 26
  4683.4  909.72  4686.4  909.59  4698.8  908.41  4709.9  908.17  4713.3  907.91
  4756.1  906.62  4764.1  906.09  4815.4  899.16  4823.7  898.25  4825.2  897.97
  4830.7   897.8  4892.8  899.46  4950.1  892.78  4991.9   884.1  4992.9   882.1
  5007.1   882.1  5008.1   884.1  5011.7   884.1    5015  885.45  5031.4  893.12
    5235  891.11  5278.5  898.11    5307  903.73  5329.7  907.72  5346.2  909.97
  5419.5  917.97
#Mann= 3 ,-1,0
  4683.4     .15       0  4991.9    .048       0  5008.1     .13       0
Bank Sta=4991.9,5008.1
XS Rating Curve= 0 ,0
Exp/Cntr=0.3,0.1

Type RM Length L Ch R = 1 ,37497   ,500,500,500
BEGIN DESCRIPTION:
Georges Creek 75.0
END DESCRIPTION:
XS GIS Cut Line= 3
        1531625.        1103025.      1531748.38      1102678.61
        1532181.      1102315.96
#Sta/Elev= 30
  4729.6  919.74    4776  913.12  4794.7  908.55  4802.4  907.64  4828.8  903.19
  4869.1  894.95  4885.9  895.96  4888.5  895.63  4905.3  892.97    4919  891.78
  4920.8  891.52  4931.1  891.04  4962.3  891.26  4979.5  890.12  4991.9  884.21
  4992.9  882.21  5007.1  882.21  5008.1  884.21  5013.4  887.46  5025.4  890.83
  5137.2   887.4  5190.9  887.58  5321.1  891.17  5380.9  890.86  5431.3  896.21
  5493.6  906.11  5508.3  912.42  5512.4  912.96  5525.3  911.26  5564.5  917.49
#Mann= 3 ,-1,0
  4729.6     .15       0  4991.9    .048       0  5008.1     .13       0
Bank Sta=4991.9,5008.1
XS Rating Curve= 0 ,0
Exp/Cntr=0.3,0.1

Type RM Length L Ch R = 1 ,36997   ,500,500,500
BEGIN DESCRIPTION:
Georges Creek 74.0
END DESCRIPTION:
XS GIS Cut Line= 3
       1532066.9      1103265.09      1532173.53      1102932.37
      1532497.38       1102570.1
#Sta/Elev= 23
  4650.6  923.28  4686.2  919.18  4688.5  919.17  4760.9  912.92  4797.6  906.85
  4801.8  906.31  4815.1  904.07  4830.7  902.46  4874.7  896.19  4883.6  894.55
  4951.9  887.53  4956.1  887.47  4991.1  884.21  4992.2  882.21  5007.8  882.21
  5008.9  884.21  5012.8  884.21  5036.3  887.39  5223.7  888.17  5278.3   900.5
  5330.2  910.47  5352.3  913.17  5392.7  923.55
#Mann= 3 ,-1,0
  4650.6     .15       0  4991.1    .048       0  5008.9     .13       0
Bank Sta=4991.1,5008.9
XS Rating Curve= 0 ,0
Exp/Cntr=0.3,0.1

Type RM Length L Ch R = 1 ,36497   ,500,500,500
BEGIN DESCRIPTION:
Georges Creek 73.0
END DESCRIPTION:
XS GIS Cut Line= 3
      1532367.72      1103441.43      1532649.91      1103074.45
      1532678.91      1102777.56
#Sta/Elev= 18
  4646.1  908.85  4727.7  903.87  4791.1  898.28  4825.2  892.58  4860.5  888.73
  4938.9  885.02  4991.9  881.41  4992.9  879.41  5007.1  879.41  5008.1  881.41
  5018.5  888.21  5019.5  888.27  5087.7  885.35  5128.2  886.38  5150.6  886.44
  5199.2  890.33  5227.6  896.63  5286.5  911.91
#Mann= 3 ,-1,0
  4646.1     .15       0  4991.9    .048       0  5008.1     .13       0
Bank Sta=4991.9,5008.1
XS Rating Curve= 0 ,0
Exp/Cntr=0.3,0.1

Type RM Length L Ch R = 1 ,35997   ,499,499,499
BEGIN DESCRIPTION:
Georges Creek 72.0
END DESCRIPTION:
XS GIS Cut Line= 3
      1533093.83      1103845.98      1533142.46       1103148.1
      1533223.49      1102746.44
#Sta/Elev= 30
  4434.2  903.81  4445.4  902.71  4487.1   900.3  4548.3  897.82  4563.4  896.12
  4607.6  893.51    4627  893.42  4657.7  891.35  4671.5   890.7  4711.6  892.05
  4729.3  891.72  4768.5  889.18  4782.5  888.92  4827.8  885.71  4838.3  885.32
  4847.9  885.55  4869.7  884.69  4895.6   884.9  4990.3  877.94  4991.5  875.94
  5008.5  875.94  5009.7  877.94  5030.7   883.2  5087.4  886.35  5242.5  886.73
  5249.3  886.75  5281.1  882.17  5320.7  894.09  5336.7  898.37    5378  905.36
#Mann= 4 ,-1,0
  4434.2     .15       0  4990.3    .048       0  5009.7     .13       0
  5242.5      10       0
Bank Sta=4990.3,5009.7
XS Rating Curve= 0 ,0
Exp/Cntr=0.3,0.1

Type RM Length L Ch R = 1 ,35498   ,499,499,499
BEGIN DESCRIPTION:
Georges Creek 71.0
END DESCRIPTION:
XS GIS Cut Line= 3
      1533657.86      1103615.18      1533637.11      1103036.88
        1533825.        1102825.
#Sta/Elev= 29
  4596.6  900.07  4620.3  898.41  4692.1  896.99  4728.6  894.65  4735.3  894.03
  4765.1  892.09  4767.4     892  4769.1  891.98  4839.2  889.46  4845.2  888.89
  4899.7  892.03    4901  891.86  4901.8  891.74  4953.2  883.91  4990.3  877.14
  4991.5  875.14  5008.5  875.14  5009.7  877.14  5019.3  880.53  5028.9  882.63
  5088.9  883.63  5170.2  883.82  5175.1  883.83    5212  882.95  5244.4  881.37
  5279.4  878.11  5339.2  898.65  5340.6  899.06  5372.1  902.86
#Mann= 5 ,-1,0
  4596.6      10       0  4901.8     .15       0  4990.3    .048       0
  5009.7     .13       0  5170.2      10       0
Bank Sta=4990.3,5009.7
XS Rating Curve= 0 ,0
Exp/Cntr=0.3,0.1

Type RM Length L Ch R = 1 ,34999   ,502,502,502
BEGIN DESCRIPTION:
Georges Creek 70.0
END DESCRIPTION:
XS GIS Cut Line= 3
      1534096.12      1103482.92      1534145.39       1103106.9
      1534267.27      1102808.68
#Sta/Elev= 20
  4678.6  898.33    4688  897.11  4715.9  894.38  4901.5  883.32  4921.4  882.59
  4984.2   875.2  4989.5   875.2  4990.8   873.2  5009.2   873.2  5010.5   875.2
  5018.2  876.12  5057.9   877.2  5096.7   878.3  5195.4  882.72  5224.7  882.96
  5237.5  886.24  5264.4  893.83  5280.1  897.19  5302.7  899.14  5313.3  898.92
#Mann= 3 ,-1,0
  4678.6    .135       0  4989.5    .048       0  5010.5    .135       0
Bank Sta=4989.5,5010.5
XS Rating Curve= 0 ,0
Exp/Cntr=0.3,0.1

Type RM Length L Ch R = 1 ,34497   ,500,500,500
BEGIN DESCRIPTION:
Georges Creek 69.0
END DESCRIPTION:
XS GIS Cut Line= 3
      1534365.82      1103545.16      1534595.81      1103289.47
      1534863.72      1103060.22
#Sta/Elev= 18
  4665.1  897.45  4706.8  893.71    4732  890.51  4793.9  884.18  4840.5  880.42
  4975.4  875.47  4991.9   875.2  4992.9   873.2  5007.1   873.2  5008.1   875.2
  5048.6   881.1  5054.6  881.14    5075  880.81  5208.3  888.78  5221.5  889.19
  5226.9  889.46  5287.3  893.63    5290  893.71
#Mann= 3 ,-1,0
  4665.1     .15       0  4991.9     .05       0  5008.1     .15       0
Bank Sta=4991.9,5008.1
XS Rating Curve= 0 ,0
Exp/Cntr=0.3,0.1

Type RM Length L Ch R = 1 ,33997   ,588,588,588
BEGIN DESCRIPTION:
Georges Creek 68.0
END DESCRIPTION:
XS GIS Cut Line= 3
      1534845.57      1103973.05      1534979.23      1103605.36
      1535203.44       1103451.8
#Sta/Elev= 11
  4629.7  896.09  4797.6  882.41  4811.5  881.61  4991.1  872.24  4992.2  870.24
  5007.8  870.24  5008.9  872.24  5025.2  873.22  5051.6  872.24  5194.6  884.65
  5271.8  894.72
#Mann= 3 ,-1,0
  4629.7     .15       0  4991.1     .05       0  5008.9     .15       0
Bank Sta=4991.1,5008.9
XS Rating Curve= 0 ,0
Exp/Cntr=0.3,0.1

Type RM Length L Ch R = 1 ,33409   ,412,412,412
BEGIN DESCRIPTION:
Georges Creek 67.0
END DESCRIPTION:
XS GIS Cut Line= 3
      1535312.36      1104356.85      1535403.12      1104017.13
      1535569.09      1103807.08
#Sta/Elev= 28
  4639.1  900.06  4640.6  900.08    4641  900.03  4641.2  900.02  4642.4  899.87
  4650.4  899.48  4682.7  896.31  4697.4  894.06  4708.6  890.56  4742.4  887.37
  4769.9  885.72    4778   884.5  4813.5  881.85  4816.8   881.5  4916.1  875.41
  4920.3  875.05  4928.8  874.92    4937  874.28  4959.1  873.48  4991.1  871.78
  4992.2  869.78  5007.8  869.78  5008.9  871.78  5018.4  872.33  5092.3  881.95
  5121.9  885.19  5150.9  892.26  5226.8   904.7
#Mann= 3 ,-1,0
  4639.1     .15       0  4991.1     .05       0  5008.9     .15       0
Bank Sta=4991.1,5008.9
XS Rating Curve= 0 ,0
Exp/Cntr=0.3,0.1

Type RM Length L Ch R = 1 ,32997   ,500,500,500
BEGIN DESCRIPTION:
Georges Creek 66.0
END DESCRIPTION:
XS GIS Cut Line= 3
      1535776.55      1104502.07      1535820.27      1104090.84
      1535820.63      1103869.32
#Sta/Elev= 19
  4616.3  893.57  4627.9  893.09  4681.4     890  4707.4  890.14  4721.5   889.1
    4732  888.67  4754.3  885.64  4802.7  875.96  4808.2  873.06  4825.5  871.12
  4925.1  875.06  4987.9  869.46  4989.4  867.46  5010.7  867.46  5012.2  869.46
    5037  873.06  5084.8  878.47  5109.5  885.46  5145.5  894.32
#Mann= 3 ,-1,0
  4616.3     .15       0  4987.9     .05       0  5012.2     .15       0
Bank Sta=4987.9,5012.2
XS Rating Curve= 0 ,0
Exp/Cntr=0.3,0.1

Type RM Length L Ch R = 1 ,32497   ,500,500,500
BEGIN DESCRIPTION:
Georges Creek 65.0
END DESCRIPTION:
XS GIS Cut Line= 3
      1536269.27      1104540.97      1536310.29      1104060.34
      1536264.08      1103820.05
#Sta/Elev= 18
  4517.6  891.65  4529.7  890.43  4533.1  889.98  4558.7  889.87  4606.5  885.29
  4651.3  883.19  4662.5  882.06  4722.2  878.37  4742.4  876.66  4823.1  871.94
  4880.3  872.34  4940.6  874.26  4987.9  868.85  4989.4  866.85  5010.7  866.85
  5012.2  868.85  5058.9  877.14  5117.7  893.23
#Mann= 3 ,-1,0
  4517.6     .15       0  4987.9     .05       0  5012.2     .15       0
Bank Sta=4987.9,5012.2
XS Rating Curve= 0 ,0
Exp/Cntr=0.3,0.1

Type RM Length L Ch R = 1 ,31997   ,467,467,467
BEGIN DESCRIPTION:
Georges Creek 64.0
END DESCRIPTION:
XS GIS Cut Line= 3
      1536761.99      1104577.28      1536803.05      1104118.22
      1536881.28      1103892.66
#Sta/Elev= 16
  4663.6  888.89  4680.2  887.94  4716.3  877.76  4727.8  875.08  4756.6  870.58
  4784.1  869.95  4905.5  873.82  4962.6  868.01  4990.3  868.01  4991.5  866.01
  5008.5  866.01  5009.7  868.01  5138.3     877  5172.3     880  5216.7   885.9
  5238.7  889.82
#Mann= 3 ,-1,0
  4663.6     .15       0  4990.3     .05       0  5009.7     .15       0
Bank Sta=4990.3,5009.7
XS Rating Curve= 0 ,0
Exp/Cntr=0.3,0.1

Type RM Length L Ch R = 1 ,31530   ,431,431,431
BEGIN DESCRIPTION:
Georges Creek 63.0
END DESCRIPTION:
XS GIS Cut Line= 3
      1537080.96      1104748.43      1537189.87      1104349.07
      1537386.96      1103980.83
#Sta/Elev= 24
  4623.2  889.24  4625.6  888.63  4687.1  874.31  4768.7  869.56  4774.6  869.05
  4784.7  868.63  4889.9  868.35  4903.9   869.3  4967.4  868.93  4972.3  868.68
  4987.1  867.86  4991.1  866.76  4992.2  864.76  5007.8  864.76  5008.9  866.76
  5040.3  871.78  5115.8  870.19    5142  868.04  5158.9  868.77  5210.9  868.93
  5295.6  874.32    5365  883.67  5388.8   888.2    5390  888.47
#Mann= 3 ,-1,0
  4623.2     .15       0  4991.1     .05       0  5008.9     .15       0
Bank Sta=4991.1,5008.9
XS Rating Curve= 0 ,0
Exp/Cntr=0.5,0.3

Type RM Length L Ch R = 1 ,31099   ,108,108,108
BEGIN DESCRIPTION:
Georges Creek 62.5
END DESCRIPTION:
XS GIS Cut Line= 4
      1537511.44      1104787.33      1537558.12      1104582.46
      1537617.76      1104432.05      1537685.18      1104203.85
#Sta/Elev= 22
  4739.7  877.59  4749.8   876.4  4756.6  876.12  4764.7  875.29  4788.5  874.47
  4794.3  874.16  4821.3  873.92  4821.9   873.9  4847.4  873.58  4906.5  870.16
  4949.8  870.84  4958.1  871.08  4988.1   868.3  4989.9   863.8  5010.2   863.8
  5011.9   868.3  5028.4  868.68  5054.3  873.59  5063.2  873.68    5135  877.34
    5163   878.1  5349.6  877.52
#Mann= 3 ,-1,0
  4739.7    .145       0  4988.1    .043       0  5011.9    .145       0
#XS Ineff= 2 , 0
          4921.5   879.4  5078.5          876.01
Permanent Ineff=
       F       F
Bank Sta=4988.1,5011.9
XS Rating Curve= 0 ,0
Exp/Cntr=0.5,0.3

Type RM Length L Ch R = 3 ,31032   ,,,
BEGIN DESCRIPTION:
Lenhardt Rd. (Georges Cr.) - TOR
Structure ID: LDS_GC_10
Approximate Survey Structure
END DESCRIPTION:
Bridge Culvert--1,0,-1,-1, 0
Deck Dist Width WeirC Skew NumUp NumDn MinLoCord MaxHiCord MaxSubmerge Is_Ogee
53.5,27,3,0, 23, 23, , , , 0, 1,1,,
    4734  4738.8  4818.9  4847.2  4854.7    4919  4932.4    4975    4975    5025
    5025  5170.1  5173.3  5176.3  5185.2  5214.7  5222.4  5224.9  5230.9  5243.2
  5245.6  5307.6    5363
  889.33  889.07  882.07  881.31  880.95  879.58   878.6     875     875     875
     875  877.74   877.9     878  877.71  877.89  878.23  878.14  878.15  878.13
  878.04  878.18  880.22
   843.8   843.8   843.8   843.8   843.8   843.8   843.8   843.8   873.5   873.5
   843.8   843.8   843.8   843.8   843.8   843.8   843.8   843.8   843.8   843.8
   843.8   843.8   843.8
    4734  4738.8  4818.9  4847.2  4854.7    4919  4932.4    4975    4975    5025
    5025  5170.1  5173.3  5176.3  5185.2  5214.7  5222.4  5224.9  5230.9  5243.2
  5245.6  5307.6    5363
  889.33  889.07  882.07  881.31  880.95  879.58   878.6     875     875     875
     875  877.74   877.9     878  877.71  877.89  878.23  878.14  878.15  878.13
  878.04  878.18  880.22
   843.8   843.8   843.8   843.8   843.8   843.8   843.8   843.8   873.5   873.5
   843.8   843.8   843.8   843.8   843.8   843.8   843.8   843.8   843.8   843.8
   843.8   843.8   843.8
Abutment Skew #Up #Dn= , 2 , 2
    4975    4976
   873.5  868.34
    4975    4976
   873.5   869.7
Abutment Skew #Up #Dn= , 2 , 2
    5024    5025
  869.26   873.5
    5024    5025
  869.02   873.5
BR Coef=-1 ,-1 , 0 ,1.25, 0 ,,,0.8,0,2,0,
WSPro=,,,, 1 ,,,, 0 ,,,, 0 ,,,,-1 ,-1 ,-1 , 0 , 0 , 0 , 0 , 0
BC Design=,, 0 ,, 0 ,,,,,,
BC HTab HWMax=878.1
BC Use User HTab Curves=0
BC User HTab FreeFlow(D)= 0

Type RM Length L Ch R = 1 ,30991   ,266,266,266
BEGIN DESCRIPTION:
Georges Creek 62.0
END DESCRIPTION:
XS GIS Cut Line= 5
      1537635.91      1104808.08      1537685.18      1104538.38
      1537695.56      1104457.99      1537752.61      1104325.73
      1537858.93      1104196.07
#Sta/Elev= 30
  4729.9  893.77  4749.1  892.62    4766   891.2  4803.5  890.41  4809.6  889.38
  4850.5  880.09  4878.5  878.74  4924.8  873.33  4932.2  872.74  4953.9  871.75
  4965.7  871.75  4980.1  868.89  4989.8  868.05  4991.4  863.55  5008.8  863.55
  5010.2  868.05  5034.1  872.14  5042.7  872.42  5082.2  872.57  5096.3  873.28
  5230.4  872.67  5249.8   872.8  5257.5  873.36  5265.7  872.79  5286.1  873.87
  5304.4  875.25  5315.4  875.49  5338.4  877.76  5360.6   879.3  5396.8  880.39
#Mann= 3 ,-1,0
  4729.9    .135       0  4989.8    .043       0  5010.2    .135       0
#XS Ineff= 2 , 0
          4947.5  877.43  5052.5          875.52
Permanent Ineff=
       F       F
Bank Sta=4989.8,5010.2
XS Rating Curve= 0 ,0
Exp/Cntr=0.5,0.3

Type RM Length L Ch R = 1 ,30725   ,200,200,200
BEGIN DESCRIPTION:
Georges Creek 61.5
END DESCRIPTION:
XS GIS Cut Line= 4
      1537717.64      1104827.58      1537843.69      1104698.07
      1537997.38      1104618.64      1538102.71      1104611.73
#Sta/Elev= 30
  4752.3  894.47  4758.7  893.67  4767.4  893.13  4773.7  892.89  4786.7   890.6
  4799.8  889.34  4814.3  887.56  4820.6   886.1  4842.3  883.03  4872.4  877.85
  4921.2  870.88  4972.4  870.66  4979.4  868.76  4991.9  862.76  4992.9  860.76
  5007.1  860.76  5008.1  862.76  5016.4  867.68  5022.8  869.25  5025.3  869.78
  5025.8  869.96    5039  870.27  5059.3  870.05  5111.1   870.5  5118.5  870.66
  5129.9  870.71  5152.9  877.51  5171.4   882.3  5193.7   890.4  5211.6  892.68
#Mann= 3 ,-1,0
  4752.3     .13       0  4991.9    .042       0  5008.1     .13       0
Bank Sta=4991.9,5008.1
XS Rating Curve= 0 ,0
Exp/Cntr=0.5,0.3

Type RM Length L Ch R = 1 ,30525   ,51,51,51
BEGIN DESCRIPTION:
Georges Creek 61.0
END DESCRIPTION:
XS GIS Cut Line= 3
      1537836.79      1104908.74      1537964.57      1104870.75
      1538179.25      1104683.78
#Sta/Elev= 19
  4814.2   884.9  4817.5  884.44  4833.3   881.4  4908.3  871.35  4947.5  870.34
  4983.3  869.56  4995.2   866.4  4997.1   860.9    5003   860.9  5004.9   866.4
  5015.2  869.41    5050  873.34  5102.4  877.71  5123.6  883.95  5141.2  887.39
  5145.5   887.6  5220.6  897.23  5226.8  898.63  5232.2  899.41
#Mann= 3 ,-1,0
  4814.2     .11       0  4995.2    .041       0  5004.9     .11       0
#XS Ineff= 2 , 0
          4982.8   870.4  5017.3           870.4
Permanent Ineff=
       F       F
Bank Sta=4995.2,5004.9
XS Rating Curve= 0 ,0
Exp/Cntr=0.5,0.3

Type RM Length L Ch R = 2 ,30505   ,,,
BEGIN DESCRIPTION:
Unnamed Trail (Georges Cr.) - TOR
Structure ID: Unnamed Trail (Georges Cr.)
Approximate Survey Structure
END DESCRIPTION:
Bridge Culvert--1,0,-1,-1, 0
Deck Dist Width WeirC Skew NumUp NumDn MinLoCord MaxHiCord MaxSubmerge Is_Ogee
15,10,3,0, 15, 15, , , , 0, 1,1,,
  4796.9  4814.4  4818.5  4893.1  4928.1  5028.5  5035.4  5076.7  5101.5  5111.5
  5139.1  5145.8  5204.1  5214.1  5227.3
  885.07  882.59  881.81  871.35   870.4   870.4  871.83  876.45   878.5  881.46
  886.85  887.18  894.67  896.92  898.82
   840.9   840.9   840.9   840.9   840.9   840.9   840.9   840.9   840.9   840.9
   840.9   840.9   840.9   840.9   840.9
  4796.9  4814.4  4818.5  4893.1  4928.1  5028.5  5035.4  5076.7  5101.5  5111.5
  5139.1  5145.8  5204.1  5214.1  5227.3
  885.07  882.59  881.81  871.35   870.4   870.4  871.83  876.45   878.5  881.46
  886.85  887.18  894.67  896.92  898.82
  840.85  840.85  840.85  840.85  840.85  840.85  840.85  840.85  840.85  840.85
  840.85  840.85  840.85  840.85  840.85
Culvert=1,4.5,4.5,10,0.015,0.4,1,1,3,860.9,5000,860.85,5000,Culvert #1  , 0 ,15
    5000    5000
BC Culvert Barrel=1,,0
Culvert Bottom n=0.015
BC Design=,, 0 ,, 0 ,,,,,,
BC HTab HWMax=899.41
BC Use User HTab Curves=0
BC User HTab FreeFlow(D)= 0

Type RM Length L Ch R = 1 ,30474   ,474,474,474
BEGIN DESCRIPTION:
Georges Creek 60.5
END DESCRIPTION:
XS GIS Cut Line= 3
      1537848.87      1104955.36      1538006.01      1104901.83
       1538204.6      1104717.06
#Sta/Elev= 25
  4780.3  884.21    4788  883.14  4797.2  880.55  4804.1   877.9  4855.5  871.62
  4926.9  869.25  4927.3  869.25  4937.4  868.79  4946.3  868.67  4978.4  868.15
  4995.2  866.35  4997.1  860.85    5003  860.85  5004.9  866.35  5023.7  868.56
    5064  876.33  5091.4  879.37  5094.1   879.5  5096.3  879.95  5097.5  880.26
  5127.7  886.17  5137.3  886.66  5175.7  891.62  5190.4  894.91  5217.5  898.82
#Mann= 3 ,-1,0
  4780.3     .11       0  4995.2    .042       0  5004.9     .11       0
#XS Ineff= 2 , 0
          4971.8   870.4  5028.3           870.4
Permanent Ineff=
       F       F
Bank Sta=4995.2,5004.9
XS Rating Curve= 0 ,0
Exp/Cntr=0.5,0.3

Type RM Length L Ch R = 1 ,30000   ,500,500,500
BEGIN DESCRIPTION:
Georges Creek 60.0
END DESCRIPTION:
XS GIS Cut Line= 3
      1538022.63      1105433.68      1538451.72      1105108.31
      1538621.79      1104920.12
#Sta/Elev= 19
  4461.5  880.88  4481.6  881.06  4565.1  875.91  4568.2  875.96  4622.2  874.05
  4667.7  869.57    4723  866.03  4889.9  868.61  4954.5  867.83  4976.7  863.19
  4991.1  860.03  4992.2  858.03  5007.8  858.03  5008.9  860.03  5030.5  867.65
  5059.8   870.7  5097.1  870.78  5136.2  877.84  5173.5  885.89
#Mann= 3 ,-1,0
  4461.5    .145       0  4991.1    .043       0  5008.9    .145       0
Bank Sta=4991.1,5008.9
XS Rating Curve= 0 ,0
Exp/Cntr=0.3,0.1

Type RM Length L Ch R = 1 ,29500   ,500,500,500
BEGIN DESCRIPTION:
Georges Creek 59.0
END DESCRIPTION:
XS GIS Cut Line= 3
        1538225.        1106025.      1538831.23      1105427.39
        1539025.        1105225.
#Sta/Elev= 30
  4352.8  873.17  4391.3  870.48  4453.9  867.28  4492.7  867.66  4500.3  867.99
  4564.3  865.69  4653.8  866.96  4691.7  864.53  4831.4  864.99  4947.5  862.24
  4985.6  859.23  4989.5  859.23  4990.8  857.23  5009.2  857.23  5010.5  859.23
  5032.6  859.34  5062.6  860.61  5068.1  861.24  5099.8  862.44  5108.8  863.82
  5114.5  863.97  5121.6  865.41  5127.6  865.59  5135.2  866.46  5151.9  866.93
  5154.9  868.07  5165.7  869.42  5183.2  872.36  5202.4  872.69  5209.6  873.97
#Mann= 3 ,-1,0
  4352.8    .145       0  4989.5    .043       0  5010.5    .145       0
Bank Sta=4989.5,5010.5
XS Rating Curve= 0 ,0
Exp/Cntr=0.3,0.1

Type RM Length L Ch R = 1 ,29000   ,458,458,458
BEGIN DESCRIPTION:
Georges Creek 58.0
END DESCRIPTION:
XS GIS Cut Line= 3
      1538679.77       1106071.5      1539160.68       1105802.5
      1539314.82      1105621.44
#Sta/Elev= 14
    4449  881.62  4585.7  868.38  4705.1  865.67  4724.3  866.38    4869  867.86
  4991.1     859  4992.2     857  5007.8     857  5008.9     859  5020.2  860.17
  5093.8  863.94    5127  866.46  5190.9  874.93  5237.8  890.01
#Mann= 3 ,-1,0
    4449    .145       0  4991.1    .043       0  5008.9    .145       0
Bank Sta=4991.1,5008.9
XS Rating Curve= 0 ,0
Exp/Cntr=0.3,0.1

Type RM Length L Ch R = 1 ,28542   ,525,525,525
BEGIN DESCRIPTION:
Georges Creek 57.0
END DESCRIPTION:
XS GIS Cut Line= 3
      1538707.38      1106231.64      1539400.42      1106192.99
      1539764.88      1105908.59
#Sta/Elev= 26
    4319  883.84  4420.6  875.19  4470.2  872.49  4608.7  860.67  4678.8  862.56
  4684.6  862.91  4968.9  860.77  4991.1  858.89  4992.2  856.89  5007.8  856.89
  5008.9  858.89  5013.2  861.72  5021.3  864.31  5047.7  863.43  5051.9  863.63
  5060.4  863.71  5091.4   865.6  5100.4  865.84  5108.6  866.23  5131.8  868.31
  5206.5  872.97  5210.6  873.14  5222.3  873.23  5329.8  879.73    5397  882.43
  5414.5  884.18
#Mann= 3 ,-1,0
    4319    .145       0  4991.1    .043       0  5008.9    .145       0
Bank Sta=4991.1,5008.9
XS Rating Curve= 0 ,0
Exp/Cntr=0.3,0.1

Type RM Length L Ch R = 1 ,28017   ,517,517,517
BEGIN DESCRIPTION:
Georges Creek 56.0
END DESCRIPTION:
XS GIS Cut Line= 4
      1539071.85      1106460.82       1539309.3      1106651.33
      1539513.62      1106723.12      1539853.24      1106524.32
#Sta/Elev= 30
  4390.5  874.05  4410.3  873.22  4459.7  874.08  4490.6  874.22    4528  872.47
  4535.9  871.57  4557.1  871.28  4570.9  870.28  4620.9  869.69  4639.7  869.86
  4674.6  868.57  4689.8  867.33  4699.7  867.07  4717.9   865.6  4728.6  865.06
  4736.1  863.91  4745.8  863.15    4759  862.82  4765.8  862.21  4828.4   860.8
  4911.5  861.54  4950.8  861.18  4991.9  858.89  4992.9  856.89  5007.1  856.89
  5008.1  858.89  5017.6  860.79  5028.9  862.03  5081.5  863.56  5225.2  877.38
#Mann= 3 ,-1,0
  4390.5    .145       0  4991.9    .043       0  5008.1    .145       0
Bank Sta=4991.9,5008.1
XS Rating Curve= 0 ,0
Exp/Cntr=0.3,0.1

Type RM Length L Ch R = 1 ,27500   ,500,500,500
BEGIN DESCRIPTION:
Georges Creek 55.0
END DESCRIPTION:
XS GIS Cut Line= 3
        1539425.        1107625.      1539839.49      1107081.36
        1540025.        1106825.
#Sta/Elev= 27
  4378.4  879.05  4415.1  875.34    4417  875.05  4432.2   873.1  4432.3   873.1
  4434.9  872.79  4437.3  872.61  4441.9  872.05    4498  866.43  4505.7  865.27
  4520.2  862.66  4571.8  864.39  4572.8  864.45  4573.7  864.55  4576.3  864.61
  4957.9  860.03  4985.5   855.7    4987   852.7    5013   852.7  5014.5   855.7
  5055.4  857.93  5078.6  857.54  5111.5  861.91  5163.6  860.68  5164.2   860.7
  5306.6  879.05  5310.2  879.44
#Mann= 3 ,-1,0
  4378.4    .145       0  4985.5    .043       0  5014.5    .145       0
Bank Sta=4985.5,5014.5
XS Rating Curve= 0 ,0
Exp/Cntr=0.3,0.1

Type RM Length L Ch R = 1 ,27000   ,521,521,521
BEGIN DESCRIPTION:
Georges Creek 54.0
END DESCRIPTION:
XS GIS Cut Line= 3
      1540328.15      1107587.35      1540337.08      1107121.87
      1540325.39      1106886.03
#Sta/Elev= 30
  4534.4  878.69  4542.1  878.07  4547.3  877.06  4553.2  875.46  4560.8  875.35
  4572.3  874.34  4575.7  874.28  4664.1  866.01  4751.2   859.5  4762.3  859.15
  4765.2   858.9  4767.8  858.39  4770.3  858.21  4782.2  858.13    4901  859.43
  4951.8  858.44  4973.7  859.35    4975  859.67    4979  858.77  4982.7  857.25
  4985.5  852.96    4987  849.96    5013  849.96  5014.5  852.96  5017.7  859.07
  5020.8   860.2  5083.6  863.58  5092.2  864.94  5101.2  867.53  5139.9  877.69
#Mann= 3 ,-1,0
  4534.4    .145       0  4985.5    .043       0  5014.5    .145       0
Bank Sta=4985.5,5014.5
XS Rating Curve= 0 ,0
Exp/Cntr=0.3,0.1

Type RM Length L Ch R = 1 ,26479   ,213,213,213
BEGIN DESCRIPTION:
Georges Creek 53.0
END DESCRIPTION:
XS GIS Cut Line= 3
      1540844.48      1107037.89      1540756.12       1106916.4
      1540620.83      1106858.42
#Sta/Elev= 17
  4854.7  873.72  4858.1  873.08  4862.8  872.56  4872.1  872.07  4888.2  870.82
  4955.2  862.04  4962.4  861.26  4968.2  860.89  4968.3  860.85  4977.8  858.25
  4979.3  857.79  4985.5     850    4987     847    5013     847  5014.5     850
  5040.4  858.84  5126.5  873.46
#Mann= 3 ,-1,0
  4854.7    .145       0  4985.5    .043       0  5014.5    .145       0
Bank Sta=4985.5,5014.5
XS Rating Curve= 0 ,0
Exp/Cntr=0.5,0.3

Type RM Length L Ch R = 1 ,26266   ,75,75,75
BEGIN DESCRIPTION:
Georges Creek 52.5
END DESCRIPTION:
XS GIS Cut Line= 4
       1541012.9      1106874.98      1540838.95      1106725.88
      1540761.64      1106665.14      1540696.16      1106610.43
#Sta/Elev= 29
    4773  868.12  4777.3  867.95  4789.8  867.82  4804.6  867.07  4811.6  865.89
  4822.1  865.36  4832.5  865.52  4836.2  865.38  4862.6  865.07  4868.5  864.63
  4876.3  864.44  4881.2  864.03  4929.2  863.53  4936.5   863.3  4949.3  863.17
  4958.4  861.81  4967.2  859.97  4968.6  860.09  4980.9  855.06  4983.6   854.3
  4988.6   847.3  5011.4   847.3  5016.6   854.3  5026.9  858.95  5035.5  860.87
  5049.8  861.37  5121.7  869.55  5168.2  873.29  5185.7  875.29
#Mann= 3 ,-1,0
    4773     .14       0  4983.6    .045       0  5016.6     .14       0
#XS Ineff= 2 , 0
          4959.5  865.75  5040.5           864.3
Permanent Ineff=
       F       F
Bank Sta=4983.6,5016.6
XS Rating Curve= 0 ,0
Exp/Cntr=0.5,0.3
