HEC-RAS study GeorgesCreek.prj: Georges Creek Limited Detail Study

--- GeorgesCreek.g06 (geometry) --- (continued)

Type RM Length L Ch R = 3 ,26239   ,,,
BEGIN DESCRIPTION:
Norman Dr. (Georges Cr.) - TOR
Structure ID: LDS_GC_09
Approximate Survey Structure
END DESCRIPTION:
Bridge Culvert--1,0,-1,-1, 0
Deck Dist Width WeirC Skew NumUp NumDn MinLoCord MaxHiCord MaxSubmerge Is_Ogee
13,28,3,0, 19, 19, , , , 0, 1,1,,
  4730.4  4820.9  4821.2  4862.8  4958.1    4961    4964  4972.5  4972.5  5027.5
  5027.5  5051.7  5054.2  5102.8    5107  5118.6  5200.3  5215.1  5216.7
  871.81  868.52  868.49  866.97  865.76  865.73   864.3   864.3   864.3   864.3
   864.3   864.3  864.91  866.93  867.52  868.03  871.16  872.06  872.05
   827.3   827.3   827.3   827.3   827.3   827.3   827.3   827.3   864.3   864.3
   827.3   827.3   827.3   827.3   827.3   827.3   827.3   827.3   827.3
  4730.4  4820.9  4821.2  4862.8  4958.1    4961    4964  4972.5  4972.5  5027.5
  5027.5  5051.7  5054.2  5102.8    5107  5118.6  5200.3  5215.1  5216.7
  871.81  868.52  868.49  866.97  865.76  865.73   864.3   864.3   864.3   864.3
   864.3   864.3  864.91  866.93  867.52  868.03  871.16  872.06  872.05
   827.3   827.3   827.3   827.3   827.3   827.3   827.3   827.3   864.3   864.3
   827.3   827.3   827.3   827.3   827.3   827.3   827.3   827.3   827.3
Abutment Skew #Up #Dn= , 2 , 2
  4972.5  4974.5
   864.3  857.68
  4972.5  4974.5
   864.3  856.78
Abutment Skew #Up #Dn= , 2 , 2
  5025.5  5027.5
  859.09   864.3
  5025.5  5027.5
  857.65   864.3
BR Coef=-1 ,-1 , 0 ,1.25, 0 ,,,0.8,0,2,0,
WSPro=,,,, 1 ,,,, 0 ,,,, 0 ,,,,-1 ,-1 ,-1 , 0 , 0 , 0 , 0 , 0
BC Design=,, 0 ,, 0 ,,,,,,
BC HTab HWMax=875.29
BC Use User HTab Curves=0
BC User HTab FreeFlow(D)= 0

Type RM Length L Ch R = 1 ,26191   ,689,689,689
BEGIN DESCRIPTION:
Georges Creek 52.0
END DESCRIPTION:
XS GIS Cut Line= 4
      1541090.77      1106838.05      1540946.04      1106715.58
       1540834.7      1106631.46      1540741.93      1106534.98
#Sta/Elev= 30
  4751.6  869.46  4768.4  868.06  4796.8  866.96  4802.4  866.47  4831.2  865.51
  4841.7  864.66    4848  864.42  4851.7   864.4  4860.5  865.11  4878.2  865.98
  4886.9  866.71  4901.8  865.06  4925.8  860.42  4930.9  859.95  4935.2  858.91
    4940  857.98  4946.8  857.82  4964.2  858.75  4974.9   856.7  4980.2  854.59
  4983.6  854.05  4988.6  847.05  5011.4  847.05  5016.6  854.05  5053.3  862.81
  5080.7  863.81  5124.7  864.87  5140.4  866.34  5189.4  869.63  5214.6     870
#Mann= 3 ,-1,0
  4751.6     .14       0  4983.6    .045       0  5016.6     .14       0
#XS Ineff= 2 , 0
          4938.5  866.01  5061.5          865.21
Permanent Ineff=
       F       F
Bank Sta=4983.6,5016.6
XS Rating Curve= 0 ,0
Exp/Cntr=0.5,0.3

Type RM Length L Ch R = 1 ,25502   ,496,496,496
BEGIN DESCRIPTION:
Georges Creek 51.0
END DESCRIPTION:
XS GIS Cut Line= 3
      1541341.48      1106192.99       1540999.1      1106013.52
        1540625.        1106025.
#Sta/Elev= 21
  4597.4  886.64  4709.4  868.04  4807.2  856.05    4899  857.27  4912.1  857.15
  4943.2   857.9  4958.7  857.36  4971.7  856.67  4980.5  854.42  4985.5  847.09
    4987  844.09    5013  844.09  5014.5  847.09  5068.2  860.43  5170.4  862.34
  5189.1   865.1  5196.5   866.5    5312  884.13  5325.8  885.26  5332.2  885.51
    5333  885.56
#Mann= 3 ,-1,0
  4597.4     .14       0  4985.5    .045       0  5014.5     .14       0
Bank Sta=4985.5,5014.5
XS Rating Curve= 0 ,0
Exp/Cntr=0.3,0.1

Type RM Length L Ch R = 1 ,25006   ,501,501,501
BEGIN DESCRIPTION:
Georges Creek 50.0
END DESCRIPTION:
XS GIS Cut Line= 4
        1541425.        1106025.      1541126.11      1105582.78
      1540974.25      1105508.23      1540645.68      1105535.85
#Sta/Elev= 30
  4431.7  876.11  4502.1  856.04  4612.2  856.18  4692.1  858.69  4730.9   858.8
  4823.7  855.47  4887.6  856.55  4941.9  853.52  4971.2   852.8  4985.5  846.05
    4987  843.05    5013  843.05  5014.5  846.05  5026.6   856.9  5030.6  858.49
    5080  857.63    5111  857.75  5261.3  859.01    5291  863.43  5296.1  864.07
  5299.1  864.85  5301.6  864.91  5325.5  868.37  5330.2  868.78  5334.3  869.03
  5339.2  870.31  5343.6  870.43  5349.8  871.34  5357.8  872.19  5416.4  880.98
#Mann= 3 ,-1,0
  4431.7     .14       0  4985.5    .045       0  5014.5     .13       0
Bank Sta=4985.5,5014.5
XS Rating Curve= 0 ,0
Exp/Cntr=0.3,0.1

Type RM Length L Ch R = 1 ,24505   ,567,567,567
BEGIN DESCRIPTION:
Georges Creek 49.0
END DESCRIPTION:
XS GIS Cut Line= 4
      1541617.59      1105861.66      1541429.83      1105486.15
      1541498.86      1105279.06      1541766.69      1105143.77
#Sta/Elev= 28
  4522.3  872.65  4523.9  872.04  4524.8  871.98  4543.2  864.96  4557.4  863.68
  4606.9  856.41  4639.6   856.5  4702.9  854.93  4709.1  855.03  4713.7  855.27
  4893.7  856.41    4905  855.91  4968.9   852.8  4985.5   845.1    4987   842.1
    5013   842.1  5014.5   845.1    5022  856.33  5023.4  856.37  5092.4  855.23
  5096.9  855.29  5108.1  855.07  5116.6  854.62  5123.3  854.57  5208.9  854.94
  5220.2  855.89  5257.2  860.26  5391.3  875.35
#Mann= 3 ,-1,0
  4522.3     .14       0  4985.5    .045       0  5014.5     .13       0
Bank Sta=4985.5,5014.5
XS Rating Curve= 0 ,0
Exp/Cntr=0.3,0.1

Type RM Length L Ch R = 1 ,23938   ,438,438,438
BEGIN DESCRIPTION:
Georges Creek 48.0
END DESCRIPTION:
XS GIS Cut Line= 4
      1542147.72       1105759.5        1541844.      1105643.53
      1541780.49      1105566.22      1541777.73      1105254.21
#Sta/Elev= 24
  4621.8  868.66  4664.7  867.11  4737.7  867.38  4811.9  861.89  4902.5  856.02
  4942.4  855.59  4946.9  854.68  4985.5  843.52    4987  840.52    5013  840.52
  5014.5  843.52  5022.1  848.52  5032.3  850.42  5046.9  850.02  5068.1  849.67
  5129.7   854.9  5165.6  856.31  5188.4  860.35  5190.9  860.56  5193.5  860.85
  5253.9  869.72  5256.1  870.13  5258.8  870.39  5262.5     871
#Mann= 3 ,-1,0
  4621.8     .15       0  4985.5    .045       0  5014.5    .135       0
Bank Sta=4985.5,5014.5
XS Rating Curve= 0 ,0
Exp/Cntr=0.3,0.1

Type RM Length L Ch R = 1 ,23500   ,500,500,500
BEGIN DESCRIPTION:
Georges Creek 47.0
END DESCRIPTION:
XS GIS Cut Line= 3
      1542236.07       1105361.9      1542049.68      1105247.53
      1541846.76      1105201.75
#Sta/Elev= 10
    4811   871.8    4884  862.92    4975   853.6  4983.1  851.03  4985.5   843.5
    4987   840.5    5013   840.5  5014.5   843.5  5037.1  850.42    5208  871.29
#Mann= 3 ,-1,0
    4811     .14       0  4985.5    .045       0  5014.5     .14       0
Bank Sta=4985.5,5014.5
XS Rating Curve= 0 ,0
Exp/Cntr=0.3,0.1

Type RM Length L Ch R = 1 ,23000   ,500,500,500
BEGIN DESCRIPTION:
Georges Creek 46.0
END DESCRIPTION:
XS GIS Cut Line= 3
      1542476.29      1105016.76      1542353.54      1104859.02
      1542175.33      1104671.62
#Sta/Elev= 14
  4800.1  875.96  4838.6  872.67  4862.2  869.82  4897.5  863.74    4948  853.29
  4983.3  847.26  4985.5   843.5    4987   840.5    5013   840.5  5014.5   843.5
  5081.4  850.42    5181  867.07  5235.8  874.05  5258.6  877.76
#Mann= 3 ,-1,0
  4800.1     .14       0  4985.5    .045       0  5014.5     .14       0
Bank Sta=4985.5,5014.5
XS Rating Curve= 0 ,0
Exp/Cntr=0.3,0.1

Type RM Length L Ch R = 1 ,22500   ,500,500,500
BEGIN DESCRIPTION:
Georges Creek 45.0
END DESCRIPTION:
XS GIS Cut Line= 3
      1542804.86      1104503.19      1542584.69      1104474.16
      1542225.03      1104436.93
#Sta/Elev= 22
  4777.9  872.77  4791.5  870.99  4791.9  871.01  4845.4  861.52  4846.7  861.38
  4928.3  854.56  4978.1   843.5  4980.7  843.73  4985.5   843.5    4987   840.5
    5013   840.5  5014.5   843.5    5042  848.93  5043.6  849.43  5072.5  854.97
  5141.7  860.57  5172.7  864.14  5182.8  865.06  5186.6  865.31  5197.1  866.96
  5214.9  870.59  5222.8   871.8
#Mann= 3 ,-1,0
  4777.9     .14       0  4985.5    .045       0  5014.5     .14       0
Bank Sta=4985.5,5014.5
XS Rating Curve= 0 ,0
Exp/Cntr=0.3,0.1

Type RM Length L Ch R = 1 ,22000   ,501,501,501
BEGIN DESCRIPTION:
Georges Creek 44.0
END DESCRIPTION:
XS GIS Cut Line= 3
      1543075.45      1104158.05      1542697.28      1103992.93
      1542410.02      1103881.94
#Sta/Elev= 30
  4593.8  881.33  4689.4  863.91  4748.1  857.71  4770.5  854.55  4777.6  853.25
  4789.5  851.41  4814.2  850.61    4858  850.41  4870.9  850.17  4880.1  849.87
  4883.2  849.94  4891.4   849.7  4959.6  852.64  4960.5  852.56  4965.4  852.79
  4985.5  843.27    4987  840.27    5013  840.27  5014.5  843.27  5059.2  848.93
  5096.9  849.56  5127.9  852.05  5208.2  861.21  5211.8  862.06  5216.9  862.58
  5219.2  863.23  5254.7  866.28  5267.9  866.15  5283.5  866.78    5308  870.53
#Mann= 3 ,-1,0
  4593.8     .14       0  4985.5    .045       0  5014.5     .14       0
Bank Sta=4985.5,5014.5
XS Rating Curve= 0 ,0
Exp/Cntr=0.3,0.1

Type RM Length L Ch R = 1 ,21499   ,520,520,520
BEGIN DESCRIPTION:
Georges Creek 43.0
END DESCRIPTION:
XS GIS Cut Line= 4
      1543180.37      1104072.46      1543078.21      1103680.38
      1543022.99       1103622.4      1542981.57      1103451.21
#Sta/Elev= 21
  4537.6  879.53  4594.6  861.13    4610  859.12  4690.6  851.85  4825.4  848.44
  4832.4  848.43  4842.3  848.18  4930.5  848.92  4946.4   849.1  4975.9  843.27
  4976.7  843.27  4985.5  843.27    4987  840.27    5013  840.27  5014.5  843.27
  5096.4  849.62  5119.9  855.15  5150.6  860.87  5162.4  865.47  5181.9  870.14
  5186.7  870.97
#Mann= 3 ,-1,0
  4537.6     .14       0  4985.5    .045       0  5014.5     .14       0
Bank Sta=4985.5,5014.5
XS Rating Curve= 0 ,0
Exp/Cntr=0.3,0.1

Type RM Length L Ch R = 1 ,20979   ,578,578,578
BEGIN DESCRIPTION:
Georges Creek 42.0
END DESCRIPTION:
XS GIS Cut Line= 4
      1543500.66      1103343.53      1543238.36      1103260.69
        1543150.      1103291.07      1542967.77      1103382.18
#Sta/Elev= 20
  4681.9  870.38  4696.8  866.74  4711.4  862.33  4809.4  856.93  4819.8  854.91
  4831.7  853.52  4847.3  852.31  4897.5  846.89  4935.9  847.93  4952.5  848.76
  4985.5  843.27    4987  840.27    5013  840.27  5014.5  843.27  5022.1  843.27
  5029.3  843.52  5065.9  845.13  5123.3  860.88  5157.7  866.53  5174.6  869.83
#Mann= 3 ,-1,0
  4681.9     .14       0  4985.5    .045       0  5014.5     .14       0
Bank Sta=4985.5,5014.5
XS Rating Curve= 0 ,0
Exp/Cntr=0.3,0.1

Type RM Length L Ch R = 1 ,20401   ,401,401,401
BEGIN DESCRIPTION:
Georges Creek 41.0
END DESCRIPTION:
XS GIS Cut Line= 3
      1543666.33       1103274.5      1543594.54      1103053.61
        1543425.        1102825.
#Sta/Elev= 15
  4841.5  863.44  4843.2  863.22    4931  848.64  4985.5   842.7    4987   839.7
    5013   839.7  5014.5   842.7    5060   852.5  5076.6   854.7  5080.3  855.29
  5098.3  857.23  5108.4  857.48  5168.8  861.67  5171.4  861.67  5233.6  865.87
#Mann= 3 ,-1,0
  4841.5     .14       0  4985.5    .045       0  5014.5     .14       0
Bank Sta=4985.5,5014.5
XS Rating Curve= 0 ,0
Exp/Cntr=0.3,0.1

Type RM Length L Ch R = 1 ,20000   ,224,224,224
BEGIN DESCRIPTION:
Georges Creek 40.0
END DESCRIPTION:
XS GIS Cut Line= 3
      1544196.46      1103039.81      1543918.93      1102856.43
      1543550.36      1102672.58
#Sta/Elev= 30
  4764.8  874.97  4792.5  873.12    4804  872.69  4806.3  872.34  4832.2  869.65
  4854.8  865.58  4870.8  863.42  4876.7  860.77  4880.8  859.79  4923.7  852.88
  4937.8  848.23  4942.7  847.49  4943.4  848.49  4959.5  845.43  4985.5  842.19
    4987  839.19    5013  839.19  5014.5  842.19  5031.8  847.49  5036.2  847.69
  5048.9   848.7  5112.1  849.36  5167.6  848.71  5238.2  849.97  5296.3  855.42
  5313.5  858.38  5321.1  859.52  5363.8  866.85  5400.7   870.1  5411.9  871.38
#Mann= 3 ,-1,0
  4764.8     .14       0  4985.5    .045       0  5014.5     .14       0
Bank Sta=4985.5,5014.5
XS Rating Curve= 0 ,0
Exp/Cntr=0.5,0.3

Type RM Length L Ch R = 1 ,19776   ,125,125,125
BEGIN DESCRIPTION:
Georges Creek 39.9
END DESCRIPTION:
XS GIS Cut Line= 4
       1544180.9      1102851.99      1544029.03      1102662.86
      1543920.04      1102613.45      1543658.46      1102565.49
#Sta/Elev= 25
  4719.4  873.92    4728  873.54  4755.1  870.33  4760.6     870  4778.2  869.32
  4840.7  862.35    4962  850.24  4975.4   846.4  4977.8   838.3  5022.2   838.3
  5024.6   846.4  5047.8  845.92  5054.6  847.01  5077.2  846.92  5079.7  847.44
  5081.6  847.44    5105  847.18  5136.5  847.59  5177.1  848.97  5186.5  849.05
  5195.8  848.72  5232.2   851.3    5246  851.68  5263.4  852.93  5347.6  860.65
#Mann= 3 ,-1,0
  4719.4     .13       0  4975.4    .043       0  5024.6     .15       0
#XS Ineff= 2 , 0
            4913  858.53    5087          853.65
Permanent Ineff=
       F       F
Bank Sta=4975.4,5024.6
XS Rating Curve= 0 ,0
Exp/Cntr=0.5,0.3

Type RM Length L Ch R = 3 ,19730   ,,,
BEGIN DESCRIPTION:
Saluda Dam Rd. - TOR
Structure ID: LDS_GC_08
Approximate Survey Structure
END DESCRIPTION:
Bridge Culvert--1,0,-1,-1, 0
Deck Dist Width WeirC Skew NumUp NumDn MinLoCord MaxHiCord MaxSubmerge Is_Ogee
27,38,3,0, 13, 13, , , , 0, 1,1,,
  4727.3    4745  4763.9  4879.7    4894  4895.4    4940    4940    5060    5060
  5193.1  5195.4  5271.7
   873.8  873.13  873.07  865.42   862.6  862.33   852.7   852.7   852.7   852.7
  857.37  857.28   858.5
   818.3   818.3   818.3   818.3   818.3   818.3   818.3   851.7   851.7   818.3
   818.3   818.3   818.3
  4727.3    4745  4763.9  4879.7    4894  4895.4    4940    4940    5060    5060
  5193.1  5195.4  5271.7
   873.8  873.13  873.07  865.42   862.6  862.33   852.7   852.7   852.7   852.7
  857.37  857.28   858.5
   818.3   818.3   818.3   818.3   818.3   818.3   818.3   851.7   851.7   818.3
   818.3   818.3   818.3
Pier Skew, UpSta & Num, DnSta & Num=  ,4970, 2 ,4970, 2 , 0 , 0 , 0 ,0,0
       1       1
  850.77   851.7
       1       1
   839.9   851.7
Pier Skew, UpSta & Num, DnSta & Num=  ,5030, 2 ,5030, 2 , 0 , 0 , 0 ,0,0
       1       1
  849.49   851.7
       1       1
  848.87   851.7
Abutment Skew #Up #Dn= , 2 , 2
    4940    4941
   851.7  854.79
    4940    4941
   851.7  844.04
Abutment Skew #Up #Dn= , 2 , 2
    5059    5060
  846.99   851.7
    5059    5060
  846.33   851.7
BR Coef=-1 ,-1 , 0 ,1.25, 0 ,,,0.8,0,2,0,
WSPro=,,,, 1 ,,,, 0 ,,,, 0 ,,,,-1 ,-1 ,-1 , 0 , 0 , 0 , 0 , 0
BC Design=,, 0 ,, 0 ,,,,,,
BC HTab HWMax=873.92
BC Use User HTab Curves=0
BC User HTab FreeFlow(D)= 0

Type RM Length L Ch R = 1 ,19651   ,89,89,89
BEGIN DESCRIPTION:
Georges Creek 39.6
END DESCRIPTION:
XS GIS Cut Line= 5
      1544216.64      1102750.74       1544127.3      1102643.53
      1544029.02      1102536.32      1543939.68      1102473.78
       1543802.7      1102420.18
#Sta/Elev= 29
  4691.5  874.22  4695.4  873.21  4741.2  869.79  4757.9  869.37    4789  867.42
  4817.4  861.41  4823.5   861.2  4842.9   859.7  4856.9  859.41  4892.6  854.28
  4954.3  841.22  4956.8  841.17  4959.3   841.3  4973.4  846.15    4976  838.05
  5024.1  838.05  5026.7  846.15  5043.6   845.6  5054.2   846.4  5085.5  845.97
  5097.6  846.11  5101.2  846.67  5120.2  850.71  5153.7  854.88  5157.5  855.42
  5168.6  855.95  5199.8  856.68  5222.4  858.32  5232.6  858.33
#Mann= 3 ,-1,0
  4691.5     .15       0  4973.4    .045       0  5026.7     .15       0
#XS Ineff= 2 , 0
            4880  865.36    5120          854.81
Permanent Ineff=
       F       F
Bank Sta=4973.4,5026.7
XS Rating Curve= 0 ,0
Exp/Cntr=0.5,0.3

Type RM Length L Ch R = 1 ,19562   ,65,65,65
BEGIN DESCRIPTION:
Georges Creek 39.3
END DESCRIPTION:
XS GIS Cut Line= 6
      1544201.75      1102381.47      1544106.45      1102384.44
      1544023.07      1102420.18      1543972.44      1102449.96
      1543886.08      1102446.98      1543784.83      1102381.47
#Sta/Elev= 27
  4782.6  863.11  4834.8   861.9  4841.4  861.28  4863.8  861.03  4869.5  860.21
  4871.4   859.9    4878   858.6  4902.3  854.43    4974  850.15  4978.3   844.8
  4980.2   838.1  5019.8   838.1  5021.8   844.8  5027.4  846.82  5056.5  849.66
  5080.8   851.2  5087.8  852.35  5113.8  854.42  5117.2  854.93    5148  855.62
  5171.3  857.22  5176.2  857.23  5187.6  858.12  5205.8  857.89  5215.7   858.8
  5232.8  861.29  5234.4  861.45
#Mann= 3 ,-1,0
  4782.6     .14       0  4978.3    .043       0  5021.8     .14       0
#XS Ineff= 2 , 0
            4954  853.42    5046           853.2
Permanent Ineff=
       F       F
Bank Sta=4978.3,5021.8
XS Rating Curve= 0 ,0
Exp/Cntr=0.5,0.3

Type RM Length L Ch R = 3 ,19532   ,,,
BEGIN DESCRIPTION:
Old Saluda Dam Rd. - TOR
Structure ID: LDS_GC_07
Approximate Survey Structure
END DESCRIPTION:
Bridge Culvert--1,0,-1,-1, 0
Deck Dist Width WeirC Skew NumUp NumDn MinLoCord MaxHiCord MaxSubmerge Is_Ogee
16,28,3,0, 25, 25, , , , 0, 1,1,,
  4754.1  4789.1  4801.4  4810.2  4816.6  4865.8  4907.7  4911.1  4950.4  4953.3
    4970    4970    5030    5030  5068.1  5075.3  5099.7  5105.3  5107.5  5133.2
  5153.3  5154.6  5160.4  5212.1  5221.5
   861.8  859.05  858.29  857.51  857.47   855.9  854.62  854.62  853.66  853.48
     852     852     852     852  852.46  853.64  854.04  855.06  855.16  857.18
  858.34  858.32  859.11  863.78  865.16
   818.1   818.1   818.1   818.1   818.1   818.1   818.1   818.1   818.1   818.1
   818.1   850.5   850.5   818.1   818.1   818.1   818.1   818.1   818.1   818.1
   818.1   818.1   818.1   818.1   818.1
  4754.1  4789.1  4801.4  4810.2  4816.6  4865.8  4907.7  4911.1  4950.4  4953.3
    4970    4970    5030    5030  5068.1  5075.3  5099.7  5105.3  5107.5  5133.2
  5153.3  5154.6  5160.4  5212.1  5221.5
   861.8  859.05  858.29  857.51  857.47   855.9  854.62  854.62  853.66  853.48
     852     852     852     852  852.46  853.64  854.04  855.06  855.16  857.18
  858.34  858.32  859.11  863.78  865.16
   818.1   818.1   818.1   818.1   818.1   818.1   818.1   818.1   818.1   818.1
   818.1   850.5   850.5   818.1   818.1   818.1   818.1   818.1   818.1   818.1
   818.1   818.1   818.1   818.1   818.1
Pier Skew, UpSta & Num, DnSta & Num=  ,5000, 2 ,5000, 2 , 0 , 0 , 0 ,0,0
       1       1
   838.1   850.5
       1       1
  837.85   850.5
Abutment Skew #Up #Dn= , 2 , 2
    4970    4971
   850.5  852.14
    4970    4971
   850.5  846.04
Abutment Skew #Up #Dn= , 2 , 2
    5029    5030
  846.98   850.5
    5029    5030
  844.37   850.5
BR Coef=-1 ,-1 , 0 ,1.25, 0 ,,,0.8,0,2,0,
WSPro=,,,, 1 ,,,, 0 ,,,, 0 ,,,,-1 ,-1 ,-1 , 0 , 0 , 0 , 0 , 0
BC Design=,, 0 ,, 0 ,,,,,,
BC HTab HWMax=863.11
BC Use User HTab Curves=0
BC User HTab FreeFlow(D)= 0

Type RM Length L Ch R = 1 ,19497   ,496,496,496
BEGIN DESCRIPTION:
Georges Creek 39.0
END DESCRIPTION:
XS GIS Cut Line= 6
      1544213.59      1102354.77      1544155.46      1102302.46
      1544092.97      1102285.02       1543992.7      1102372.21
      1543868.21      1102372.53      1543778.87      1102309.99
#Sta/Elev= 30
  4716.1   858.6  4717.4  858.49  4747.7  859.02  4757.5  858.96  4765.1  857.88
  4779.9   855.5  4794.3  852.85  4804.7  851.66    4833  846.68  4835.6  846.36
  4839.4  845.53  4847.2  844.29  4859.2  840.81  4862.1  840.46  4868.5  840.72
  4879.7  837.48    4918  837.74  4938.5  838.37  4976.4  844.18  4978.4  837.48
  5021.6  837.48  5023.8  844.18  5041.7  844.12  5080.8  850.11  5095.6  853.02
  5112.2  858.42  5122.3  858.26  5206.9  869.87  5214.8  870.68  5225.6  871.32
#Mann= 3 ,-1,0
  4716.1     .14       0  4976.4    .043       0  5023.8     .14       0
#XS Ineff= 2 , 0
            4949  853.69    5051          853.03
Permanent Ineff=
       F       F
Bank Sta=4976.4,5023.8
XS Rating Curve= 0 ,0
Exp/Cntr=0.5,0.3

Type RM Length L Ch R = 1 ,19001   ,516,516,516
BEGIN DESCRIPTION:
Georges Creek 38.0
END DESCRIPTION:
XS GIS Cut Line= 3
      1544355.12      1102411.25      1544355.12      1102107.49
        1544225.        1101825.
#Sta/Elev= 26
  4606.2  863.24  4619.9  860.45  4641.2  860.49  4708.6  843.46  4740.3  837.93
  4747.9  836.95  4770.5  837.24  4776.9  837.14  4808.3  837.69  4830.4  837.39
  4863.6  838.11  4879.9  837.48  4896.6  837.35    4910  836.68  4935.3  835.33
  4947.8   832.4  4953.9  831.31  4985.4  824.77  4985.5   824.6    4987   821.6
    5013   821.6  5014.5   824.6  5031.7   824.6    5088  842.95  5220.5  874.09
    5221  874.22
#Mann= 3 ,-1,0
  4606.2     .14       0  4985.5    .043       0  5014.5     .14       0
Bank Sta=4985.5,5014.5
XS Rating Curve= 0 ,0
Exp/Cntr=0.3,0.1

Type RM Length L Ch R = 1 ,18485   ,503,503,503
BEGIN DESCRIPTION:
Georges Creek 37.0
END DESCRIPTION:
XS GIS Cut Line= 4
      1544897.11      1102113.45      1544825.64      1101964.55
      1544718.43      1101881.16      1544444.46      1101791.82
#Sta/Elev= 19
  4798.7  860.47  4916.2  837.19  4927.7   835.8  4953.9  824.94    4955  824.58
  4967.4   819.5  4985.5  819.45    4987  816.45    5013  816.45  5014.5  819.45
  5053.4  832.16    5060  832.58  5090.9  833.35    5150  835.65  5233.3  836.03
    5237  836.34  5328.3  850.62  5339.3   852.7  5358.1  856.94
#Mann= 3 ,-1,0
  4798.7     .14       0  4985.5    .043       0  5014.5     .14       0
Bank Sta=4985.5,5014.5
XS Rating Curve= 0 ,0
Exp/Cntr=0.3,0.1

Type RM Length L Ch R = 1 ,17982   ,482,482,482
BEGIN DESCRIPTION:
Georges Creek 36.0
END DESCRIPTION:
XS GIS Cut Line= 3
        1545025.        1101425.      1544712.48      1101529.76
      1544456.37      1101505.94
#Sta/Elev= 13
  4841.6  847.05  4905.1  830.87  4915.3  828.65  4954.3  818.28  4958.1  817.45
  4985.5  817.45    4987  814.45    5013  814.45  5014.5  817.45  5022.7  830.32
  5171.2  833.21  5254.5  833.51  5414.1  865.24
#Mann= 3 ,-1,0
  4841.6     .14       0  4985.5    .043       0  5014.5     .14       0
Bank Sta=4985.5,5014.5
XS Rating Curve= 0 ,0
Exp/Cntr=0.3,0.1

Type RM Length L Ch R = 1 ,17500   ,500,500,500
BEGIN DESCRIPTION:
Georges Creek 35.0
END DESCRIPTION:
XS GIS Cut Line= 3
        1545025.        1101025.      1544736.45      1101027.88
        1544625.        1101025.
#Sta/Elev= 19
  4711.4   863.5  4801.8  854.22  4812.8  851.75  4817.8   849.9  4856.4  841.34
  4863.8  840.22    4957  829.02  4959.2  828.65  4960.3  828.29  4985.5  817.34
    4987  814.34  4999.9  814.34  5000.1  814.34    5013  814.34  5014.5  817.34
  5026.6  817.34  5046.5  830.89  5066.2  839.68  5111.5  855.53
#Mann= 3 ,-1,0
  4711.4     .14       0  4999.9    .043       0  5000.1     .14       0
Bank Sta=4985.5,5014.5
XS Rating Curve= 0 ,0
Exp/Cntr=0.3,0.1

Type RM Length L Ch R = 1 ,17000   ,500,500,500
BEGIN DESCRIPTION:
Georges Creek 34.0
END DESCRIPTION:
XS GIS Cut Line= 3
        1545225.        1101025.      1545036.37      1100746.39
        1544825.        1100625.
#Sta/Elev= 20
  4663.5  870.44  4709.5  870.39  4827.4  858.77  4883.9  844.45  4924.2  832.64
  4949.8  828.51  4968.3  817.23  4969.8  815.95  4982.3  815.95  4983.8  812.95
  5016.2  812.95  5017.7  815.95  5036.1   828.3  5044.5  833.12  5071.3   832.9
  5089.7  834.98  5129.1  840.85  5190.9  868.33  5194.3   870.2  5199.1  871.87
#Mann= 3 ,-1,0
  4663.5     .14       0  4982.3    .042       0  5017.7     .14       0
Bank Sta=4982.3,5017.7
XS Rating Curve= 0 ,0
Exp/Cntr=0.3,0.1

Type RM Length L Ch R = 1 ,16500   ,500,500,500
BEGIN DESCRIPTION:
Georges Creek 33.0
END DESCRIPTION:
XS GIS Cut Line= 3
        1545425.        1100625.      1545404.27      1100422.07
        1545225.        1100225.
#Sta/Elev= 18
    4796  837.21  4829.5  829.86  4848.1  829.86  4897.3  828.65  4919.7  824.88
  4968.4   818.7  4982.3  815.72  4983.8  812.72  5016.2  812.72  5017.7  815.72
  5031.4  815.72  5043.4  819.38  5073.2  830.35  5146.5  832.51  5147.1  832.66
  5208.7  845.75  5210.2  846.19  5210.7   846.4
#Mann= 3 ,-1,0
    4796     .14       0  4982.3    .042       0  5017.7     .14       0
Bank Sta=4982.3,5017.7
XS Rating Curve= 0 ,0
Exp/Cntr=0.3,0.1

Type RM Length L Ch R = 1 ,16000   ,500,500,500
BEGIN DESCRIPTION:
Georges Creek 32.0
END DESCRIPTION:
XS GIS Cut Line= 3
        1546225.        1100425.      1545684.36      1100051.27
        1545625.        1099825.
#Sta/Elev= 23
  4374.7  847.76  4463.3  829.38  4554.5   829.7  4558.4   830.6  4659.3  831.65
  4853.6  829.52  4926.1  830.49  4941.3  825.38  4954.8  820.33  4977.1  815.38
  4982.3  815.38  4983.8  812.38  5016.2  812.38  5017.7  815.38  5037.9  815.38
  5059.5  830.04  5065.1  833.51  5084.5  836.16  5089.7  837.11  5102.4  838.88
  5107.6  839.33  5109.8  839.99  5143.1  848.27
#Mann= 3 ,-1,0
  4374.7     .14       0  4982.3    .042       0  5017.7     .14       0
Bank Sta=4982.3,5017.7
XS Rating Curve= 0 ,0
Exp/Cntr=0.3,0.1

Type RM Length L Ch R = 1 ,15500   ,500,500,500
BEGIN DESCRIPTION:
Georges Creek 31.0
END DESCRIPTION:
XS GIS Cut Line= 3
        1546225.        1100425.      1546174.21      1100114.21
        1546025.        1099625.
#Sta/Elev= 30
  4724.9  847.47  4801.6  834.32  4836.7  829.27  4882.6  828.12  4898.4  827.28
  4932.9  820.27    4939  819.63  4963.3  816.69    4972  815.38  4982.3  815.38
  4983.8  812.38  5016.2  812.38  5017.7  815.38  5051.2  815.38  5081.9  820.38
  5150.7  824.18  5233.8  826.68  5242.6   827.6  5299.6  829.38  5301.1  829.63
  5315.8   830.9  5328.4  832.32  5348.6  833.31  5351.7  833.93  5396.9  838.49
  5436.9  839.48  5444.4  839.46  5451.6  839.66  5484.4   841.8  5511.5  842.92
#Mann= 3 ,-1,0
  4724.9     .14       0  4982.3    .042       0  5017.7     .11       0
Bank Sta=4982.3,5017.7
XS Rating Curve= 0 ,0
Exp/Cntr=0.3,0.1

Type RM Length L Ch R = 1 ,15000   ,544,544,544
BEGIN DESCRIPTION:
Georges Creek 30.0
END DESCRIPTION:
XS GIS Cut Line= 3
      1546615.84      1100053.39      1546580.56      1099907.07
      1546480.86      1099529.58
#Sta/Elev= 23
  4849.5  842.31  4863.8  842.67  4867.3  842.66  4913.7  831.02  4930.3  827.21
  4948.7  820.17  4957.5  813.72  4982.3  813.71  4983.8  810.71  5016.2  810.71
  5017.7  813.71  5019.4  817.59    5021  818.03  5092.7   818.1  5101.6  819.67
  5130.6  827.65    5158  827.11  5206.3   827.3  5275.6  829.04  5275.9  829.05
  5287.2  829.41  5339.7  829.02  5390.4  836.54
#Mann= 3 ,-1,0
  4849.5     .14       0  4982.3    .043       0  5017.7     .14       0
Bank Sta=4982.3,5017.7
XS Rating Curve= 0 ,0
Exp/Cntr=0.3,0.1

Type RM Length L Ch R = 1 ,14456   ,499,499,499
BEGIN DESCRIPTION:
Georges Creek 29.0
END DESCRIPTION:
XS GIS Cut Line= 4
      1547081.23      1099966.76      1547024.82      1099898.26
      1547024.82      1099821.71        1547025.        1099625.
#Sta/Elev= 26
  4830.3  843.72  4872.8  834.93  4879.2   834.2    4919  828.86  4922.8  828.46
  4925.8  827.91  4926.2  827.97  4928.6  826.89    4975   811.6  4975.2  811.57
  4982.3  811.57  4983.8  808.57  5016.2  808.57  5017.7  811.57  5024.1  815.49
  5036.3  820.72  5042.7  825.65  5105.4  826.97  5129.4  828.16  5134.8  828.32
  5141.8  828.68  5145.9  828.81  5146.4  828.77  5149.1   829.4  5158.6  830.11
  5192.3  834.54
#Mann= 3 ,-1,0
  4830.3     .14       0  4982.3    .043       0  5017.7     .14       0
Bank Sta=4982.3,5017.7
XS Rating Curve= 0 ,0
Exp/Cntr=0.3,0.1

Type RM Length L Ch R = 1 ,13957   ,493,493,493
BEGIN DESCRIPTION:
Georges Creek 28.0
END DESCRIPTION:
XS GIS Cut Line= 3
      1547431.79      1099555.77      1547331.05      1099465.11
      1547198.08      1099414.74
#Sta/Elev= 15
  4852.3  844.99  4877.2  838.44  4955.5  826.65  4971.6  815.98  4980.9  810.35
  4982.3  810.35  4983.8  807.35  5016.2  807.35  5017.7  810.35  5023.3  810.51
  5030.4  814.43  5044.1  822.35  5050.7  825.88  5095.6  838.52    5130  845.45
#Mann= 3 ,-1,0
  4852.3     .14       0  4982.3    .043       0  5017.7     .14       0
Bank Sta=4982.3,5017.7
XS Rating Curve= 0 ,0
Exp/Cntr=0.3,0.1

Type RM Length L Ch R = 1 ,13464   ,497,497,497
BEGIN DESCRIPTION:
Georges Creek 27.0
END DESCRIPTION:
XS GIS Cut Line= 3
        1547825.        1099425.       1547750.1      1099231.41
      1547679.59      1099094.41
#Sta/Elev= 16
  4787.7  836.03  4806.2  833.31  4861.2  828.35  4882.8  826.84  4891.8  825.57
  4947.8  824.93  4968.3  809.62  4982.3  809.62  4983.8  806.62  5016.2  806.62
  5017.7  809.62  5034.4  821.11  5053.1  828.74    5067  832.22    5113  842.06
  5149.3  848.52
#Mann= 3 ,-1,0
  4787.7     .14       0  4982.3    .043       0  5017.7     .14       0
Bank Sta=4982.3,5017.7
XS Rating Curve= 0 ,0
Exp/Cntr=0.3,0.1

Type RM Length L Ch R = 1 ,12967   ,564,564,564
BEGIN DESCRIPTION:
Georges Creek 26.0
END DESCRIPTION:
XS GIS Cut Line= 4
      1548191.32      1099382.51       1548189.3      1099207.23
      1548213.48      1099150.82      1548251.76      1099062.17
#Sta/Elev= 15
  4764.1  844.32  4795.6  838.05  4813.2  833.06  4881.1  824.71  4939.4  822.83
  4955.6  822.38  4962.8  817.72  4973.6  809.62  4982.3  809.62  4983.8  806.62
  5016.2  806.62  5017.7  809.62  5031.6  809.62  5074.3  843.17  5097.4  864.87
#Mann= 3 ,-1,0
  4764.1     .14       0  4982.3    .043       0  5017.7     .14       0
Bank Sta=4982.3,5017.7
XS Rating Curve= 0 ,0
Exp/Cntr=0.5,0.3

Type RM Length L Ch R = 1 ,12403   ,135,135,135
BEGIN DESCRIPTION:
Georges Creek 25.0
END DESCRIPTION:
XS GIS Cut Line= 4
      1548874.08      1099301.55      1548869.72      1099236.16
      1548729.24      1099166.94      1548452.64      1099089.38
#Sta/Elev= 26
  4771.3  841.02  4835.7  829.21  4836.9  829.33  4839.9  829.39  4877.2  832.63
  4932.1  824.38  4943.2  821.42  4951.8  823.66  4954.4  823.87  4984.3   819.1
    4990     807    5010     807  5015.8   819.1  5028.5  815.57  5061.4   829.4
  5107.2  839.63  5192.8  848.39  5197.1  850.89  5214.9  854.25  5219.4  855.74
  5226.9  857.56  5228.4  857.65  5237.8  862.38  5249.7  867.49  5261.6  866.91
  5280.8  869.21
#Mann= 3 ,-1,0
  4771.3     .13       0  4984.3    .042       0  5015.8     .13       0
#XS Ineff= 2 , 0
            4879  833.07    5121          847.67
Permanent Ineff=
       F       F
Bank Sta=4984.3,5015.8
XS Rating Curve= 0 ,0
Exp/Cntr=0.5,0.3

Type RM Length L Ch R = 3 ,12365   ,,,
BEGIN DESCRIPTION:
Latham Rd. (Georges Cr.) - TOR
Structure ID: LDS_GC_06
Approximate Survey Structure
END DESCRIPTION:
Bridge Culvert--1,0,-1,-1, 0
Deck Dist Width WeirC Skew NumUp NumDn MinLoCord MaxHiCord MaxSubmerge Is_Ogee
21,34,3,0, 14, 14, , , , 0, 1,1,,
  4725.5  4725.9  4748.4  4791.9  4820.6  4833.9  4886.3  4897.9    4900    4900
    5100    5100  5107.2  5321.7
  843.97  843.94  840.26  829.38  832.34  832.42  833.18  831.63   832.7   832.7
   832.7   832.7  846.82  860.01
     787     787     787     787     787     787     787     787     787   828.7
   828.7     787     787     787
  4725.5  4725.9  4748.4  4791.9  4820.6  4833.9  4886.3  4897.9    4900    4900
    5100    5100  5107.2  5321.7
  843.97  843.94  840.26  829.38  832.34  832.42  833.18  831.63   832.7   832.7
   832.7   832.7  846.82  860.01
     787     787     787     787     787     787     787     787     787   828.7
   828.7     787     787     787
Pier Skew, UpSta & Num, DnSta & Num=  ,4950, 2 ,4950, 2 , 0 , 0 , 0 ,0,0
       4       4
  823.19   828.7
       4       4
  817.34   828.7
Pier Skew, UpSta & Num, DnSta & Num=  ,5050, 2 ,5050, 2 , 0 , 0 , 0 ,0,0
       4       4
  824.61   828.7
       4       4
  824.69   828.7
Abutment Skew #Up #Dn= , 2 , 2
    4900    4910
   828.7   827.7
    4900    4910
   828.7  822.29
Abutment Skew #Up #Dn= , 2 , 2
    5090    5100
  839.88   828.7
    5090    5100
  831.64   828.7
BR Coef=-1 ,-1 , 0 ,1.25, 0 ,,,0.8,0,2,0,
WSPro=,,,, 1 ,,,, 0 ,,,, 0 ,,,,-1 ,-1 ,-1 , 0 , 0 , 0 , 0 , 0
BC Design=,, 0 ,, 0 ,,,,,,
BC HTab HWMax=869.21
BC Use User HTab Curves=0
BC User HTab FreeFlow(D)= 0

Type RM Length L Ch R = 1 ,12268   ,302,302,302
BEGIN DESCRIPTION:
Georges Creek 24.5
END DESCRIPTION:
XS GIS Cut Line= 5
      1548920.58      1099301.55      1548952.55      1099162.04
      1548872.62      1099128.62      1548807.23      1099093.74
      1548515.13        1099008.
#Sta/Elev= 30
  4742.4   844.8  4748.1  844.34  4802.4  829.49  4826.3  831.74  4847.8  831.81
  4874.7  824.43  4885.6  823.66  4947.6  820.19  4979.6  818.85    4987  806.75
    5013  806.75  5020.5  818.85  5038.7  823.04  5078.1   829.1  5084.5  830.59
  5089.4  831.36  5137.7  844.87    5142  845.43  5155.9  849.01  5172.7  854.06
  5201.2  858.07  5227.5  861.51  5237.9  862.23  5250.2  865.13  5268.9  868.08
  5278.1  869.16  5292.6  871.55  5307.6  872.45  5331.8  874.23  5350.7  877.58
#Mann= 3 ,-1,0
  4742.4     .13       0  4979.6    .042       0  5020.5     .13       0
#XS Ineff= 2 , 0
            4820  832.28    5180           851.3
Permanent Ineff=
       F       F
Bank Sta=4979.6,5020.5
XS Rating Curve= 0 ,0
Exp/Cntr=0.5,0.3

Type RM Length L Ch R = 1 ,11966   ,273,273,273
BEGIN DESCRIPTION:
Georges Creek 24.0
END DESCRIPTION:
XS GIS Cut Line= 4
      1549021.24      1099207.96      1549148.85      1099063.89
      1549109.74      1098971.28        1549025.        1098825.
#Sta/Elev= 24
    4707  829.03  4736.3  825.34  4740.5  825.47  4764.8  825.11    4776  824.38
  4807.8  823.08  4835.7  823.25  4884.1  821.71    4898  821.55  4899.5  821.56
  4904.7  821.23  4908.6  820.81  4964.2  817.06  4968.8  814.68  4978.8  808.81
  4980.6  805.81  5019.4  805.81  5021.2  808.81  5024.9  809.62  5048.7  823.71
    5088  824.29  5131.2  831.05  5149.3   833.2  5169.1  834.96
#Mann= 3 ,-1,0
    4707     .14       0  4978.8    .043       0  5021.2    .115       0
Bank Sta=4978.8,5021.2
XS Rating Curve= 0 ,0
Exp/Cntr=0.5,0.3

Type RM Length L Ch R = 1 ,11693   ,297,297,297
BEGIN DESCRIPTION:
Georges Creek 23.0
END DESCRIPTION:
XS GIS Cut Line= 4
      1549910.95      1099041.42      1549336.13      1098845.73
      1549245.38      1098808.91      1548620.49       1098625.8
#Sta/Elev= 30
  4389.1  866.84  4435.9  867.42  4700.3  830.53    4736  832.71  4811.7  833.66
  4846.8  832.53  4850.1  831.14  4877.1  828.44  4913.3  829.14  4936.2  826.01
  4951.7  820.71  4976.4  814.68  4977.5   812.1  4981.5   805.1  5018.5   805.1
  5022.5   812.1  5056.1   824.2  5104.6  822.37  5138.1   828.3    5210  836.89
  5301.3  845.62  5389.7  845.89  5415.4  848.39  5434.8  852.09  5515.8  857.69
  5580.2  865.86  5600.5  866.72  5644.1  874.03  5681.6  878.01  5745.4  881.13
#Mann= 3 ,-1,0
  4389.1    .115       0  4977.5     .04       0  5022.5    .115       0
#XS Ineff= 2 , 0
            4733  900.33    5267           900.1
Permanent Ineff=
       F       F
Bank Sta=4977.5,5022.5
XS Rating Curve= 0 ,0
Exp/Cntr=0.5,0.3

Type RM Length L Ch R = 3 ,11546   ,,,
BEGIN DESCRIPTION:
Southern Railway (Georges Cr.) - TOR
Structure ID: Southern Railway (Georges Cr.)
Approximate Survey Structure
END DESCRIPTION:
Bridge Culvert--1,0,-1,-1, 0
Deck Dist Width WeirC Skew NumUp NumDn MinLoCord MaxHiCord MaxSubmerge Is_Ogee
117,60,3,0, 29, 29, , , , 0, 1,1,,
  4264.7  4319.5    4320  4320.2  4320.3  4321.2    4463  4471.2    4472  4472.6
  4473.3    4475  4490.3  4738.7  4743.3  4743.9  4744.1  4744.4  4744.8  4745.2
  4745.5  4748.3  4767.5    4850    4850    5150    5150    5514  5688.7
  904.65   904.6  904.62  904.61  904.59  904.55  902.81  901.93  901.89   901.7
  901.64  901.52  901.93  900.29  900.16  900.07  900.07  900.06  900.02  900.04
  900.01  900.26   900.1   900.1   900.1   900.1   900.1   900.1   900.4
   785.1   785.1   785.1   785.1   785.1   785.1   785.1   785.1   785.1   785.1
   785.1   785.1   785.1   785.1   785.1   785.1   785.1   785.1   785.1   785.1
   785.1   785.1   785.1   785.1   897.1   897.1   785.1   785.1   785.1
  4264.7  4319.5    4320  4320.2  4320.3  4321.2    4463  4471.2    4472  4472.6
  4473.3    4475  4490.3  4738.7  4743.3  4743.9  4744.1  4744.4  4744.8  4745.2
  4745.5  4748.3  4767.5    4850    4850    5150    5150    5514  5688.7
  904.65   904.6  904.62  904.61  904.59  904.55  902.81  901.93  901.89   901.7
  901.64  901.52  901.93  900.29  900.16  900.07  900.07  900.06  900.02  900.04
  900.01  900.26   900.1   900.1   900.1   900.1   900.1   900.1   900.4
   785.1   785.1   785.1   785.1   785.1   785.1   785.1   785.1   785.1   785.1
   785.1   785.1   785.1   785.1   785.1   785.1   785.1   785.1   785.1   785.1
   785.1   785.1   785.1   785.1   897.1   897.1   785.1   785.1   785.1
Pier Skew, UpSta & Num, DnSta & Num=  ,4880, 2 ,4880, 2 , 0 , 0 , 0 ,0,0
       2       2
  828.37   897.1
       2       2
  822.48   897.1
Pier Skew, UpSta & Num, DnSta & Num=  ,4940, 2 ,4940, 2 , 0 , 0 , 0 ,0,0
       2       2
  824.71   897.1
       2       2
   819.7   897.1
Pier Skew, UpSta & Num, DnSta & Num=  ,5000, 2 ,5000, 2 , 0 , 0 , 0 ,0,0
       2       2
   805.1   897.1
       2       2
  804.85   897.1
Pier Skew, UpSta & Num, DnSta & Num=  ,5060, 2 ,5060, 2 , 0 , 0 , 0 ,0,0
       2       2
  824.01   897.1
       2       2
  824.19   897.1
Pier Skew, UpSta & Num, DnSta & Num=  ,5120, 2 ,5120, 2 , 0 , 0 , 0 ,0,0
       2       2
  825.17   897.1
       2       2
  830.97   897.1
Abutment Skew #Up #Dn= , 2 , 2
    4850    4900
   897.1  828.21
    4850    4900
   897.1   822.2
Abutment Skew #Up #Dn= , 2 , 2
    5100    5150
  822.45   897.1
    5100    5150
  828.83   897.1
BR Coef=-1 ,-1 , 0 ,1.25, 0 ,,,0.8,0,2,0,
WSPro=,,,, 1 ,,,, 0 ,,,, 0 ,,,,-1 ,-1 ,-1 , 0 , 0 , 0 , 0 , 0
BC Design=,, 0 ,, 0 ,,,,,,
BC HTab HWMax=881.13
BC Use User HTab Curves=0
BC User HTab FreeFlow(D)= 0

Type RM Length L Ch R = 1 ,11396   ,355,355,355
BEGIN DESCRIPTION:
Georges Creek 22.5
END DESCRIPTION:
XS GIS Cut Line= 5
      1550056.27      1098771.12      1549675.53      1098628.71
      1549474.02      1098576.13      1549283.16       1098532.8
      1548681.53      1098439.79
#Sta/Elev= 30
  4279.6  901.91  4427.2  890.25  4499.1  874.41  4547.5  866.29    4579  855.81
  4609.9  847.93  4622.1  847.82  4662.3  840.63  4700.8  831.86  4728.2  830.51
  4768.7  831.14  4785.9  826.99  4811.5  827.39  4875.9  822.56  4947.9  819.42
  4973.2  815.38  4977.5  811.85  4981.5  804.85  5018.5  804.85  5022.5  811.85
  5046.1  822.57  5234.6  843.26  5324.2  844.36  5422.5  849.97  5456.8  854.25
    5516  855.41  5545.3  859.68  5611.4  863.98    5653  869.86  5698.8  872.69
#Mann= 3 ,-1,0
  4279.6    .115       0  4977.5     .04       0  5022.5    .115       0
#XS Ineff= 2 , 0
            4730  900.35    5270           900.1
Permanent Ineff=
       F       F
Bank Sta=4977.5,5022.5
XS Rating Curve= 0 ,0
Exp/Cntr=0.5,0.3

Type RM Length L Ch R = 1 ,11041   ,546,546,546
BEGIN DESCRIPTION:
Georges Creek 22.0
END DESCRIPTION:
XS GIS Cut Line= 3
      1549783.95      1098510.01      1549641.57       1098328.8
      1549517.32       1098147.6
#Sta/Elev= 26
  4761.7  828.92  4790.2  819.67  4873.1  821.32  4958.3  817.94  4969.1  811.01
  4973.7  807.88  4979.3  807.65  4981.3  803.65  5018.7  803.65  5020.7  807.65
  5034.5  821.17  5066.4  819.67  5066.7  819.77  5068.3  819.82  5071.7  820.66
    5075  820.79  5079.2  821.11  5108.3  824.66  5122.5  825.85  5131.2  826.35
  5144.6  828.32  5150.9  829.67  5153.6  830.32  5162.4  831.14  5164.6  831.71
  5170.6  832.56
#Mann= 3 ,-1,0
  4761.7     .15       0  4979.3    .046       0  5020.7     .15       0
Bank Sta=4979.3,5020.7
XS Rating Curve= 0 ,0
Exp/Cntr=0.3,0.1

Type RM Length L Ch R = 1 ,10495   ,595,595,595
BEGIN DESCRIPTION:
Georges Creek 21.0
END DESCRIPTION:
XS GIS Cut Line= 4
      1550156.71      1098196.78      1550060.93       1097966.4
       1549908.2       1097875.8      1549664.87      1097870.62
#Sta/Elev= 25
    4647   842.7  4722.7  821.79    4726  821.39  4803.5  819.31  4868.8  821.86
    4890  820.46  4896.5  820.19  4960.7  816.32  4973.6  812.18  4979.3  807.77
  4981.3  803.77  5018.7  803.77  5020.7  807.77  5069.1  818.73  5074.1  818.47
    5079  818.26  5100.2  816.32  5102.2  816.34  5122.3  819.51    5133  820.81
    5211  833.11  5236.3  835.49  5255.7  838.72  5266.5  839.56  5304.8  843.79
#Mann= 3 ,-1,0
    4647     .15       0  4979.3    .046       0  5020.7     .15       0
Bank Sta=4979.3,5020.7
XS Rating Curve= 0 ,0
Exp/Cntr=0.3,0.1

Type RM Length L Ch R = 1 ,9900    ,438,438,438
BEGIN DESCRIPTION:
Georges Creek 20.0
END DESCRIPTION:
XS GIS Cut Line= 3
      1550607.12       1097466.8      1550236.95      1097440.91
      1549662.28      1097446.09
#Sta/Elev= 29
  4647.2  843.24  4747.2  832.38  4750.2  832.13  4768.9  831.78  4787.1  830.52
  4814.5  829.69  4831.4  828.67  4850.3  826.84  4887.6  820.11  4918.7  817.04
    4919  816.98  4919.3  816.92    4927     816    4973  809.43  4979.3   806.5
  4981.3   802.5  5018.7   802.5  5020.7   806.5  5051.8  818.98  5165.5   818.8
  5258.7  814.73  5334.8  818.07  5370.2  817.13    5419  817.13  5473.2  819.09
  5486.8  822.97  5513.1  832.28  5516.4   832.5  5568.3  841.06
#Mann= 3 ,-1,0
  4647.2     .15       0  4979.3    .046       0  5020.7     .15       0
Bank Sta=4979.3,5020.7
XS Rating Curve= 0 ,0
Exp/Cntr=0.3,0.1

Type RM Length L Ch R = 1 ,9462    ,460,460,460
BEGIN DESCRIPTION:
Georges Creek 19.0
END DESCRIPTION:
XS GIS Cut Line= 3
      1550076.46      1097021.56      1549833.13      1097223.47
      1549670.05      1097264.89
#Sta/Elev= 24
  4883.6  834.16  4898.6  830.29  4908.8  826.51    4968  816.32  4972.6  815.25
  4976.7  809.56  4979.2  805.92  4979.3  805.92  4981.3  801.92  5018.7  801.92
  5020.7  805.92    5034   806.5  5054.7  812.39  5103.6   811.7  5125.8  813.52
  5143.8  814.15  5179.3  816.22  5185.9  816.66  5201.2  817.33  5224.1  819.52
  5249.2  822.61  5301.5  827.41  5322.8  831.02  5347.6  834.22
#Mann= 3 ,-1,0
  4883.6     .15       0  4979.3    .046       0  5020.7     .15       0
Bank Sta=4979.3,5020.7
XS Rating Curve= 0 ,0
Exp/Cntr=0.3,0.1

Type RM Length L Ch R = 1 ,9002    ,502,502,502
BEGIN DESCRIPTION:
Georges Creek 18.0
END DESCRIPTION:
XS GIS Cut Line= 3
      1549776.18      1096638.44      1549659.69      1096765.28
      1549582.04      1097024.15
#Sta/Elev= 18
  4847.9  833.69  4895.6  822.87  4946.3   817.3  4953.6   816.8  4970.5  815.33
  4977.1  809.95  4979.3   805.8  4981.3   801.8  5018.7   801.8  5020.7   805.8
  5048.9  815.62  5049.6  815.86  5050.1   815.8    5100  811.29  5111.5  810.66
  5128.9  811.99  5187.8  821.33  5223.9  833.51
#Mann= 4 ,-1,0
  4847.9     .15       0  4979.3    .046       0  5020.7     .15       0
  5048.9      10       0
Bank Sta=4979.3,5020.7
XS Rating Curve= 0 ,0
Exp/Cntr=0.3,0.1

Type RM Length L Ch R = 1 ,8500    ,500,500,500
BEGIN DESCRIPTION:
Georges Creek 17.0
END DESCRIPTION:
XS GIS Cut Line= 3
      1549789.12      1096506.42      1549449.96      1096442.21
      1549286.93      1096418.41
#Sta/Elev= 28
  4673.3  844.09  4687.7  841.47  4702.2  838.43  4717.5   836.1  4756.6   832.1
  4765.4   831.4    4769  830.93  4771.6  830.31  4773.7  829.88  4839.1  819.67
  4853.2  818.14    4855  817.99  4860.4  817.42  4898.4   815.8  4931.6  815.28
  4962.9  813.78  4972.3  803.38  4979.3  803.38  4981.3  799.38  5018.7  799.38
  5020.7  803.38  5021.5  804.82  5037.2  816.95  5087.5  837.12  5092.8  838.95
  5094.6  839.51  5095.9  840.04    5104  842.65
#Mann= 3 ,-1,0
  4673.3     .15       0  4979.3    .046       0  5020.7     .15       0
Bank Sta=4979.3,5020.7
XS Rating Curve= 0 ,0
Exp/Cntr=0.3,0.1

Type RM Length L Ch R = 1 ,8000    ,522,522,522
BEGIN DESCRIPTION:
Georges Creek 16.0
END DESCRIPTION:
XS GIS Cut Line= 3
      1549970.33      1096270.86      1549728.48      1096032.43
        1549425.        1096025.
#Sta/Elev= 30
    4757  833.48  4768.8  830.91  4774.1  830.47    4782  828.31  4795.4  826.98
  4802.5  826.73  4846.6  822.04  4893.5   815.7  4914.3  814.33  4961.9  813.08
  4978.4  802.22  4979.3  802.22  4981.3  798.22  5018.7  798.22  5020.7  802.22
  5025.3  803.52  5042.4   812.5  5056.3  813.73  5075.2  814.33  5105.4  811.57
  5117.1   812.5  5157.8  817.28  5168.2  819.19  5187.9  820.22    5211  822.61
  5223.9  822.65    5250  824.59  5266.2  824.51  5276.8  825.95  5303.6  828.74
#Mann= 3 ,-1,0
    4757     .15       0  4979.3    .046       0  5020.7     .15       0
Bank Sta=4979.3,5020.7
XS Rating Curve= 0 ,0
Exp/Cntr=0.3,0.1

Type RM Length L Ch R = 1 ,7478    ,478,478,478
BEGIN DESCRIPTION:
Georges Creek 15.0
END DESCRIPTION:
XS GIS Cut Line= 3
      1550172.24      1095755.73      1550068.69      1095644.42
      1549864.19      1095571.94
#Sta/Elev= 24
  4839.2  821.81  4851.8  820.61  4862.3  818.92  4899.4  813.88    4920  811.94
  4928.3  813.43  4958.3   800.6  4979.3   800.6  4981.3   796.6  5018.7   796.6
  5020.7   800.6    5024     807  5028.8  809.78  5030.6  810.73  5035.9  812.85
  5038.5  813.29  5039.7   813.3  5041.3  813.38  5066.1  814.93  5080.2  818.78
  5084.5  819.75    5095  822.65  5108.8  824.14  5123.1  825.38
#Mann= 3 ,-1,0
  4839.2     .15       0  4979.3    .045       0  5020.7     .15       0
Bank Sta=4979.3,5020.7
XS Rating Curve= 0 ,0
Exp/Cntr=0.3,0.1

Type RM Length L Ch R = 1 ,7000    ,580,580,580
BEGIN DESCRIPTION:
Georges Creek 14.0
END DESCRIPTION:
XS GIS Cut Line= 3
        1550589.      1095675.48      1550326.46      1095246.59
      1550094.58      1095038.68
#Sta/Elev= 17
  4556.7  822.41  4605.2  816.38  4628.3  816.08  4700.4  811.87  4833.5  808.13
  4919.6  811.65  4979.3  800.26  4981.3  796.26  5018.7  796.26  5020.7  800.26
  5026.3  805.58    5040  811.19  5055.6  811.77  5088.2  812.32  5107.6  812.04
  5151.9  820.68    5260     821
#Mann= 3 ,-1,0
  4556.7     .15       0  4979.3    .042       0  5020.7     .11       0
Bank Sta=4979.3,5020.7
XS Rating Curve= 0 ,0
Exp/Cntr=0.5,0.3

Type RM Length L Ch R = 1 ,6420    ,39,39,39
BEGIN DESCRIPTION:
Georges Creek 13.0
END DESCRIPTION:
XS GIS Cut Line= 2
    1551220.9265    1095051.0574    1550283.4392    1094621.2055
#Sta/Elev= 30
  4371.5  820.81  4433.8  814.98  4495.2  811.66  4533.4  810.26  4616.9  809.07
  4632.3  808.36  4636.2  809.08  4704.6  808.97  4834.8  810.23  4898.1  808.37
  4934.9  807.95  4956.2  808.43    4960 804.386  4964.6  799.49  4966.7  796.35
  4979.9  796.17  4995.6  796.81  5002.7  799.36  5005.4  802.75  5011.2  803.51
  5029.2  802.86  5043.6  811.39  5054.6   819.6  5103.7  820.42  5126.7  820.95
  5183.9  823.12  5310.8  829.46  5363.2  836.01  5391.2  837.76  5402.8  837.94
#Mann= 3 ,-1,0
  4371.5     .15       0  4956.2    .042       0  5103.7      .1       0
#XS Ineff= 2 , 0
       0  4859.3  824.38  5111.3       0  824.38
Permanent Ineff=
       F       F
Bank Sta=4960,5005.4
XS Rating Curve= 0 ,0
Exp/Cntr=0.5,0.3

Type RM Length L Ch R = 1 ,6381    ,86,86,86
BEGIN DESCRIPTION:
Georges Creek 13.0
END DESCRIPTION:
XS GIS Cut Line= 4
    1551237.1813    1095015.6063    1551237.1813    1095015.6063
1550554.584369411094702.62543343     1550299.694    1094585.7544
#Sta/Elev= 30
 4351.75  828.24 4424.85  824.76 4514.65  821.38 4614.78  819.11  4718.6  819.34
 4820.41  820.16  4903.9  819.82 4923.91  817.79 4940.24  807.04 4942.95  805.77
 4957.47  805.61 4962.89  800.88 4970.11  798.09 4976.65  798.03 4989.56   796.1
 4993.89     796 5009.15  797.06 5018.42  804.45 5022.18  805.94 5033.51  811.83
 5041.54  813.58 5045.82  813.98 5055.89  817.76 5067.13  821.22 5073.13  822.01
  5079.6  821.67 5119.15  823.04 5238.34  828.45 5251.38  828.28 5383.09  834.78
#Mann= 3 ,-1,0
 4351.75     .15       0 4957.47    .042       0 5018.42      .1       0
#XS Ineff= 2 , 0
       0 4898.55  824.49 5072.55       0  824.49
Permanent Ineff=
       F       F
Bank Sta=4957.47,5018.42
XS Rating Curve= 0 ,0
Exp/Cntr=0.5,0.3

Type RM Length L Ch R = 3 ,6350    ,,,
BEGIN DESCRIPTION:
Old Easley Hwy. - TOR
Structure ID: LDS_GC_04
Approximate Survey Structure
END DESCRIPTION:
Bridge Culvert--1,0,-1,-1, 0
Deck Dist Width WeirC Skew NumUp NumDn MinLoCord MaxHiCord MaxSubmerge Is_Ogee
1,46.25,3,0, 43, 36, , , , 0, 1,1,,
  4399.3  4419.3  4439.3  4459.3  4479.3  4499.3  4519.3  4539.3  4559.3  4579.3
  4599.3  4619.3  4639.3  4659.3  4679.3  4699.3  4719.3  4739.3  4759.3  4779.3
  4799.3  4819.3  4839.3  4859.3  4879.3  4899.3  4899.3  5071.3  5071.3  5091.3
  5113.3  5133.3  5153.3  5173.3  5193.3  5213.3  5233.3  5253.3  5273.3  5293.3
  5313.3  5333.3  5353.3
  828.65  828.07  827.53  827.03  826.58  826.17   825.8  825.47  825.19  824.94
  824.74  824.57  824.37  824.34  824.38  824.47  824.57  824.67  824.77  824.87
  824.97  825.07  825.17  825.27  825.37  825.47  825.47   826.8   826.8  827.12
  827.48  827.88  828.33  828.81  829.34   829.9  830.51  831.16  831.85  832.58
  833.36  834.17  835.02
                                                                                
                                                                                
                                                  820.38  821.65
                                                                                
                        
  4412.2  4432.2  4452.2  4472.2  4492.2  4512.2  4532.2  4552.2  4572.2  4592.2
  4612.2  4632.2  4652.2  4672.2  4692.2  4712.2  4732.2  4752.2  4772.2  4792.2
  4812.2  4832.2  4852.2  4872.2  4892.2  4912.1  4912.1  5084.1  5084.1  5104.1
  5124.1  5144.1  5164.1  5184.1  5204.1  5224.1
  828.65  828.07  827.53  827.03  826.58  826.17   825.8  825.47  825.19  824.94
  824.74  824.57  824.37  824.34  824.38  824.47  824.57  824.67  824.77  824.87
  824.97  825.07  825.17  825.27  825.37  825.47  825.47   826.8   826.8  827.12
  827.48  827.88  828.33  828.81  829.34   829.9
                                                                                
                                                                                
                                                  820.38  821.65
                                                
Pier Skew, UpSta & Num, DnSta & Num=  ,4939.8, 2 ,4952.6, 2 , 0 , 0 , 0 ,,
       4       4
     800     824
       4       4
     800     824
Pier Skew, UpSta & Num, DnSta & Num=  ,5024.8, 2 ,5037.6, 2 , 0 , 0 , 0 ,,
       4       4
     800     824
       4       4
     800     824
Abutment Skew #Up #Dn= , 3 , 3
 4899.25 4901.25 4921.25
     817     817     807
  4912.1  4914.1  4934.1
     817     817     807
Abutment Skew #Up #Dn= , 3 , 3
  5049.3  5069.3  5071.3
  810.25  820.25  820.25
  5062.1  5082.1  5084.1
  810.25  820.25  820.25
BR Coef=-1 ,-1 , 0 ,1.25, 0 ,,,0.8,0,2,0,
WSPro=,,,, 1 ,,,, 0 ,,,, 0 ,,,,-1 ,-1 ,-1 , 0 , 0 , 0 , 0 , 0
BC Design=,, 0 ,, 0 ,,,,,,
BC HTab HWMax=843.14
BC Use User HTab Curves=0
BC User HTab FreeFlow(D)= 0
