HEC-RAS study GeorgesCreek.prj: Georges Creek Limited Detail Study

--- GeorgesCreek.g01 (geometry) --- (continued)

Type RM Length L Ch R = 1 ,405     ,67,67,67
BEGIN DESCRIPTION:
Georges Creek 1.5
END DESCRIPTION:
XS GIS Cut Line= 5
      1553658.04      1090044.52       1553533.3      1089910.98
      1553399.75      1089811.18      1553228.33      1089697.53
      1553031.41      1089701.12
#Sta/Elev= 30
  4615.1  819.18  4638.9  819.09  4658.9  818.24  4676.8  817.89  4703.2  811.18
    4711   810.7  4715.3  809.14  4736.2  805.85  4745.4  804.93  4808.5  802.77
  4812.4  802.43  4848.2  801.78  4870.4  801.02  4886.6  801.55    4909  800.81
  4929.1  799.21  4948.6   799.4  4964.6  794.92  4974.6  795.15  4982.4  783.75
  5017.8  783.75  5025.6  795.15  5062.9  799.52  5137.5  802.92    5157  802.69
  5170.3  803.61  5196.3  806.63  5301.8  815.15  5342.8     819  5367.2  820.46
#Mann= 3 ,-1,0
  4615.1     .13       0  4974.6     .04       0  5025.6     .13       0
#XS Ineff= 2 , 0
       0  4857.5  819.18  5142.5       0  819.28
Permanent Ineff=
       F       F
Bank Sta=4974.6,5025.6
XS Rating Curve= 0 ,0
Exp/Cntr=0.5,0.3

--- GeorgesCreek.g02 (geometry) ---

Geom Title=Corrected Effective
Program Version=6.10

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
River Reach=Georges Creek   ,Reach-1

Type RM Length L Ch R = 1 ,6420    ,39,39,39
BEGIN DESCRIPTION:
Georges Creek 13.0
END DESCRIPTION:
XS GIS Cut Line= 2
    1551220.9265    1095051.0574    1550283.4392    1094621.2055
#Sta/Elev= 30
  4371.5  820.81  4433.8  814.98  4495.2  811.66  4533.4  810.26  4616.9  809.07
  4632.3  808.36  4636.2  809.08  4704.6  808.97  4834.8  810.23  4898.1  808.37
  4934.9  807.95  4956.2  808.43    4960 804.386  4964.6  799.49  4966.7  796.35
  4979.9  796.17  4995.6  796.81  5002.7  799.36  5005.4  802.75  5011.2  803.51
  5029.2  802.86  5043.6  811.39  5054.6   819.6  5103.7  820.42  5126.7  820.95
  5183.9  823.12  5310.8  829.46  5363.2  836.01  5391.2  837.76  5402.8  837.94
#Mann= 3 ,-1,0
  4371.5     .15       0  4956.2    .042       0  5103.7      .1       0
Bank Sta=4960,5005.4
XS Rating Curve= 0 ,0
Exp/Cntr=0.5,0.3

Type RM Length L Ch R = 1 ,6381    ,86,86,86
BEGIN DESCRIPTION:
Georges Creek 13.0
END DESCRIPTION:
XS GIS Cut Line= 4
    1551237.1813    1095015.6063    1551237.1813    1095015.6063
1550554.584369411094702.62543343     1550299.694    1094585.7544
#Sta/Elev= 30
 4371.75  828.24 4444.85  824.76 4534.65  821.38 4634.78  819.11  4738.6  819.34
 4840.41  820.16  4923.9  819.82 4943.91  817.79 4960.24  807.04 4962.95  805.77
 4977.47  805.61 4982.89  800.88 4990.11  798.09 4996.65  798.03 5009.56   796.1
 5013.89     796 5029.15  797.06 5038.42  804.45 5042.18  805.94 5053.51  811.83
 5061.54  813.58 5065.82  813.98 5075.89  817.76 5087.13  821.22 5093.13  822.01
  5099.6  821.67 5139.15  823.04 5258.34  828.45 5271.38  828.28 5403.09  834.78
#Mann= 3 ,-1,0
 4371.75     .15       0 4977.47    .042       0 5038.42      .1       0
#XS Ineff= 2 , 0
       0  4884.8  821.51 5129.47       0  821.51
Permanent Ineff=
       F       F
Bank Sta=4977.47,5038.42
XS Rating Curve= 0 ,0
Exp/Cntr=0.5,0.3

Type RM Length L Ch R = 3 ,6315    ,,,
BEGIN DESCRIPTION:
Old Easley Hwy. - TOR
Structure ID: LDS_GC_04
Approximate Survey Structure
END DESCRIPTION:
Bridge Culvert--1,0,-1,-1, 0
Deck Dist Width WeirC Skew NumUp NumDn MinLoCord MaxHiCord MaxSubmerge Is_Ogee
38,36,3,0, 101, 101, , , , 0, 1,1,,
  4371.5 4378.964382.864  4383.24388.4614401.3384406.5864410.5254412.3794421.558
4430.0454437.1174437.8764438.4174447.9654448.7614453.8394462.2044470.3554475.687
4482.0684486.5414487.4414489.5424495.8114503.5574510.1144521.8094532.3244537.422
4540.8064541.3474550.2264559.6414591.9224605.2024617.6154633.6334644.0624644.813
 4655.424664.4944709.4794742.1454746.127 4751.74 4778.774798.7544815.0954839.658
4843.5694843.5874844.2284855.3414866.5874892.0544910.732  4922.8  4922.8 4937.47
4939.7364942.1074944.6184944.618  5077.3  5077.3 5091.47 5091.475100.2975100.725
5106.5755133.0045147.8345158.4895186.0875192.0735192.2155192.2615192.3645192.501
5192.5495192.7075210.937  5213.15239.255 5262.155281.9165292.364 5292.425292.582
5298.8485318.9895350.7345367.0135391.2875397.3595399.5415401.6355406.1855419.167
5434.951
 828.775 828.501 828.358 828.346 828.163 827.713 827.529 827.391 827.326 827.003
 826.705 826.455 826.428 826.407 826.071 826.042  825.86 825.561 825.269 825.078
 824.849 824.689 824.657 824.606 824.453 824.265 824.105  823.82 823.563 823.439
 823.359 823.346 823.186 823.017 822.436 822.197 821.973 821.683 821.491  821.49
 821.475 821.463 821.402 821.358 821.343 821.382 821.572 821.712 821.827 821.999
 822.027 822.027 822.029 822.062 822.095  822.17 822.225  822.28  822.28  822.29
  822.31 822.317 822.326 822.326  822.33  822.33  822.34  822.34 822.369 822.373
 822.554 823.372 823.831 824.161 825.016 825.201 825.206 825.208 825.212 825.219
 825.221 825.229 826.136 826.244 827.542 828.678 829.659 830.178 830.178 830.188
 830.506 831.526 833.135  833.96  835.19 835.498 835.609 835.714 835.941 836.588
 837.375
                                                                                
                                                                                
                                                                                
                                                                                
                                                                                
                                                           820.2   820.2  820.21
  820.23  820.24  820.25  820.25  820.25  820.25  820.26
                                                                                
                                                                                
                                                                                
        
  4371.5 4378.964382.864  4383.24388.4614401.3384406.5864410.5254412.3794421.558
4430.0454437.1174437.8764438.4174447.9654448.7614453.8394462.2044470.3554475.687
4482.0684486.5414487.4414489.5424495.8114503.5574510.1144521.8094532.3244537.422
4540.8064541.3474550.2264559.6414591.9224605.2024617.6154633.6334644.0624644.813
 4655.424664.4944709.4794742.1454746.127 4751.74 4778.774798.7544815.0954839.658
4843.5694843.5874844.2284855.3414866.5874892.0544910.732  4922.8  4922.8 4937.47
4939.7364942.1074944.6184944.618  5077.3  5077.3 5091.47 5091.475100.2975100.725
5106.5755133.0045147.8345158.4895186.0875192.0735192.2155192.2615192.3645192.501
5192.5495192.7075210.937  5213.15239.255 5262.155281.9165292.364 5292.425292.582
5298.8485318.9895350.7345367.0135391.2875397.3595399.5415401.6355406.1855419.167
5434.951
 828.775 828.501 828.358 828.346 828.163 827.713 827.529 827.391 827.326 827.003
 826.705 826.455 826.428 826.407 826.071 826.042  825.86 825.561 825.269 825.078
 824.849 824.689 824.657 824.606 824.453 824.265 824.105  823.82 823.563 823.439
 823.359 823.346 823.186 823.017 822.436 822.197 821.973 821.683 821.491  821.49
 821.475 821.463 821.402 821.358 821.343 821.382 821.572 821.712 821.827 821.999
 822.027 822.027 822.029 822.062 822.095  822.17 822.225  822.28  822.28  822.29
  822.31 822.317 822.326 822.326  822.33  822.33  822.34  822.34 822.369 822.373
 822.554 823.372 823.831 824.161 825.016 825.201 825.206 825.208 825.212 825.219
 825.221 825.229 826.136 826.244 827.542 828.678 829.659 830.178 830.178 830.188
 830.506 831.526 833.135  833.96  835.19 835.498 835.609 835.714 835.941 836.588
 837.375
                                                                                
                                                                                
                                                                                
                                                                                
                                                                                
                                                           820.2   820.2  820.21
  820.23  820.24  820.25  820.25  820.25  820.25  820.26
                                                                                
                                                                                
                                                                                
        
Pier Skew, UpSta & Num, DnSta & Num=  ,4944.8, 2 ,4944.8, 2 , 0 , 0 , 0 ,0,0
    1.75    1.75
  809.22   820.8
    1.75    1.75
  805.66   820.8
Pier Skew, UpSta & Num, DnSta & Num=  ,4966.8, 2 ,4966.8, 2 , 0 , 0 , 0 ,0,0
    1.75    1.75
  810.17   820.8
    1.75    1.75
  805.03   820.8
Pier Skew, UpSta & Num, DnSta & Num=  ,4988.8, 2 ,4988.8, 2 , 0 , 0 , 0 ,0,0
    1.75    1.75
   794.5   820.8
    1.75    1.75
  794.25   820.8
Pier Skew, UpSta & Num, DnSta & Num=  ,5010.8, 2 ,5010.8, 2 , 0 , 0 , 0 ,0,0
    1.75    1.75
   794.5   820.8
    1.75    1.75
  794.25   820.8
Pier Skew, UpSta & Num, DnSta & Num=  ,5032.8, 2 ,5032.8, 2 , 0 , 0 , 0 ,0,0
    1.75    1.75
   811.8   820.8
    1.75    1.75
  803.26   820.8
Pier Skew, UpSta & Num, DnSta & Num=  ,5054.8, 2 ,5054.8, 2 , 0 , 0 , 0 ,0,0
    1.75    1.75
  818.59   820.8
    1.75    1.75
  815.79   820.8
Abutment Skew #Up #Dn= , 2 , 2
  4922.8 4943.37
     820     808
  4922.8 4943.37
     820     808
Abutment Skew #Up #Dn= , 2 , 2
 5090.47 5091.47
  819.22  820.08
 5090.47 5091.47
  819.22  820.08
BR Coef=-1 ,-1 , 0 ,1.25, 0 ,,,0.8,0,2,0,
WSPro=,,,, 1 ,,,, 0 ,,,, 0 ,,,,-1 ,-1 ,-1 , 0 , 0 , 0 , 0 , 0
BC Design=,, 0 ,, 0 ,,,,,,
BC HTab HWMax=843.14
BC Use User HTab Curves=0
BC User HTab FreeFlow(D)= 0

Type RM Length L Ch R = 1 ,6295    ,75,75,75
BEGIN DESCRIPTION:
Georges Creek 13.0
END DESCRIPTION:
XS GIS Cut Line= 2
    1551273.0254    1094937.4321     1550335.538    1094507.5802
#Sta/Elev= 30
  4371.5  828.13  4444.6  824.65  4534.4  821.27 4634.53     819 4738.35  819.23
 4840.16  820.05 4923.65  819.71 4943.66  817.68 4959.99  806.93  4962.7  805.66
 4977.22   805.5 4982.64  800.77 4989.86  797.98  4996.4  797.92 5009.31  795.99
 5013.64  795.89  5028.9  796.95 5038.17  804.34 5041.93  805.83 5053.26  811.72
 5061.29  813.47 5065.57  813.87 5075.64  817.65 5086.88  821.11 5092.88   821.9
 5099.35  821.56  5138.9  822.93 5258.09  828.34 5271.13  828.17 5402.84  834.67
#Mann= 3 ,-1,0
  4371.5     .15       0 4977.22    .042       0 5038.17      .1       0
#XS Ineff= 2 , 0
       0  4904.8   821.4 5109.47       0   821.4
Permanent Ineff=
       F       F
Bank Sta=4977.22,5038.17
XS Rating Curve= 0 ,0
Exp/Cntr=0.5,0.3

Type RM Length L Ch R = 1 ,6220    ,260,260,260
XS GIS Cut Line= 2
    1551320.6064    1094872.9437    1550360.5379    1094437.7468
#Sta/Elev= 30
    4430     845    4665  844.67 4690.89  843.94 4699.84  836.89 4710.87  834.46
 4742.87   814.6 4748.83  811.77 4758.32  809.73  4785.9  808.23 4811.28  809.69
 4959.12  810.55 4963.54  809.08 4967.95  803.04 4975.67  801.63 4983.62  798.23
 5010.98  797.48  5015.4  798.64 5018.98  801.76 5022.02  806.74    5025   809.4
 5036.29  811.13  5050.7  822.32 5069.46  833.99 5078.43  832.24 5159.93  833.15
 5200.76   835.3 5242.48  839.45 5285.72  839.07 5311.09  843.73  5337.7   846.4
#Mann= 4 ,-1,0
    4430     .15       0    4665     .15       0 4975.67    .045       0
 5018.98     .12       0
#XS Ineff= 2 , 0
       0  4774.8  820.36  5225.3       0  820.36
Permanent Ineff=
       F       F
Bank Sta=4975.67,5018.98
XS Rating Curve= 0 ,0
Exp/Cntr(USF)=0,0
Exp/Cntr=0.5,0.3

Type RM Length L Ch R = 1 ,5800    ,42,42,42
BEGIN DESCRIPTION:
Georges Creek 11.5
END DESCRIPTION:
XS GIS Cut Line= 2
      1551170.49       1094192.6    1550419.6349    1094182.1911
#Sta/Elev= 30
    4603  825.18    4603  825.16  4608.2  822.06    4613  820.71  4657.6  817.26
    4683  818.22  4708.6  814.43  4780.6  811.83  4792.1  811.52  4832.7  812.66
  4907.8  808.45  4966.9  807.99  4974.5  803.83  4982.9  797.01    4993  797.36
  5001.3   796.6  5016.6  796.52  5023.5  797.02  5031.6   804.9  5035.6  809.22
  5083.5  811.55  5090.9  813.53  5101.4  812.92  5126.7  830.04  5144.9  837.21
  5273.9  840.19  5282.4  841.34  5339.4  844.16  5348.8  845.35  5353.9  848.08
#Mann= 3 ,-1,0
    4603     .13       0  4974.5     .04       0  5031.6      .1       0
#XS Ineff= 2 , 0
       0    4816  834.26    5184       0   837.8
Permanent Ineff=
       F       F
Bank Sta=4974.5,5031.6
XS Rating Curve= 0 ,0
Exp/Cntr=0.5,0.3

Type RM Length L Ch R = 1 ,5758    ,127,127,127
BEGIN DESCRIPTION:
Georges Creek 11.5
END DESCRIPTION:
XS GIS Cut Line= 2
    1551171.0722     1094150.604     1550420.217    1094140.1951
#Sta/Elev= 30
    4603  832.37 4606.91  832.37 4618.43  826.94 4630.42  825.06 4681.53  823.56
 4701.16  820.84 4730.48  819.92 4766.87  823.82 4790.84  823.76 4868.79  820.39
 4881.33  818.91 4894.71  814.58 4906.78  808.31 4968.19  807.45  4974.5  803.62
 4985.11  796.37 5006.02  796.03 5020.42   796.4  5031.6  805.75  5038.1     810
  5053.6  812.12 5086.16  821.84 5136.57  823.65 5159.13  830.65 5165.88  835.65
 5179.53  837.91 5227.28  837.57 5240.96  838.66 5271.01  844.59 5353.93  848.93
#Mann= 3 ,-1,0
    4603     .13       0  4974.5     .04       0  5031.6      .1       0
#XS Ineff= 2 , 0
       0    4872  834.26    5128       0  834.26
Permanent Ineff=
       F       F
Bank Sta=4974.5,5031.6
XS Rating Curve= 0 ,0
Exp/Cntr=0.5,0.3

Type RM Length L Ch R = 3 ,5677    ,,,
BEGIN DESCRIPTION:
US Hwy 123 (Georges Cr.) - TOR
Structure ID: LDS_GC_03
Approximate Survey Structure
END DESCRIPTION:
Bridge Culvert--1,0,-1,-1, 0
Deck Dist Width WeirC Skew NumUp NumDn MinLoCord MaxHiCord MaxSubmerge Is_Ogee
28,78,3,0, 20, 20, , , , 0, 1,1,,
    4603 4630.26 4630.73 4680.33 4730.12 4780.09  4830.3  4883.7    4900    4900
    5100    5100 5146.87 5196.91 5246.78 5246.78 5297.07 5297.07 5346.71 5396.73
 839.271 838.263 838.248 836.737 835.487 834.602 834.282 834.257 834.257 834.257
 837.904 837.904 839.803 842.112 844.467 844.467 846.856 846.856 849.443 851.924
                                                                           831.5
  835.14
    4603 4630.26 4630.73 4680.33 4730.12 4780.09  4830.3  4883.7    4900    4900
    5100    5100 5146.87 5196.91 5246.78 5246.78 5297.07 5297.07 5346.71 5396.73
 839.271 838.263 838.248 836.737 835.487 834.602 834.282 834.257 834.257 834.257
 837.904 837.904 839.803 842.112 844.467 844.467 846.856 846.856 849.443 851.924
                                                                           831.5
  835.14
Pier Skew, UpSta & Num, DnSta & Num=  ,4925, 2 ,4925, 2 , 0 , 0 , 0 ,0,0
    2.33    2.33
  808.63     832
    2.33    2.33
  810.79     832
Pier Skew, UpSta & Num, DnSta & Num=  ,4975, 2 ,4975, 2 , 0 , 0 , 0 ,0,0
    2.33    2.33
  805.77     833
    2.33    2.33
  805.52     833
Pier Skew, UpSta & Num, DnSta & Num=  ,5025, 2 ,5025, 2 , 0 , 0 , 0 ,0,0
    2.33    2.33
  805.77   834.6
    2.33    2.33
  805.52   834.6
Pier Skew, UpSta & Num, DnSta & Num=  ,5075, 2 ,5075, 2 , 0 , 0 , 0 ,0,0
    2.33    2.33
  809.44   835.6
    2.33    2.33
  815.52   835.6
Abutment Skew #Up #Dn= , 10 , 10
    4900 4902.39 4904.05 4907.63 4908.73 4911.98 4923.34 4925.11 4929.03 4941.87
 830.465 830.465  827.77 826.686 826.475 824.555 817.377  816.54 814.314 808.123
    4900 4902.39 4904.05 4907.63 4908.73 4911.98 4923.34 4925.11 4929.03 4941.87
 830.465 830.465  827.77 826.686 826.475 824.555 817.377  816.54 814.314 808.123
Abutment Skew #Up #Dn= , 8 , 8
    5054 5054.43 5060.64 5063.99 5072.63 5074.05 5075.51    5100
     810  811.08   816.1  818.38  823.04  823.92  824.56  833.04
    5054 5054.43 5060.64 5063.99 5072.63 5074.05 5075.51    5100
     810  811.08   816.1  818.38  823.04  823.92  824.56  833.04
BR Coef=-1 ,-1 , 0 ,1.25, 0 ,,,0.8,0,2,0,
WSPro=,,,, 1 ,,,, 0 ,,,, 0 ,,,,-1 ,-1 ,-1 , 0 , 0 , 0 , 0 , 0
BC Design=,, 0 ,, 0 ,,,,,,
BC HTab HWMax=845.29
BC Use User HTab Curves=0
BC User HTab FreeFlow(D)= 0

Type RM Length L Ch R = 1 ,5631    ,43,43,43
BEGIN DESCRIPTION:
Georges Creek 11.5
END DESCRIPTION:
XS GIS Cut Line= 2
    1551172.8326    1094023.6162    1550421.9774    1094013.2073
#Sta/Elev= 30
    4628  836.91 4654.91  835.79  4704.8  834.99 4752.48  834.99  4762.8  834.47
 4768.53  832.21 4804.86  830.19 4896.89  829.58 4911.73  826.97 4931.69  814.73
 4946.53  808.17 4956.48   805.8 4971.03  806.29 4979.42  799.29 4982.84  796.23
 5003.29  795.28  5021.2  796.46 5021.99  797.91 5024.45  799.92 5034.19  808.03
 5065.63  814.83 5102.32  833.27  5110.2  835.63 5306.74  846.23 5315.57  845.47
 5327.31  847.28 5339.32  848.04 5365.62  849.05 5372.73  848.45 5378.93  848.88
#Mann= 3 ,-1,0
    4628     .13       0 4979.42     .04       0 5024.45      .1       0
#XS Ineff= 2 , 0
       0    4891   831.5    5123       0   831.5
Permanent Ineff=
       F       F
Bank Sta=4979.42,5024.45
XS Rating Curve= 0 ,0
Exp/Cntr=0.5,0.3

Type RM Length L Ch R = 1 ,5588    ,588,588,588
BEGIN DESCRIPTION:
Georges Creek 11.0
END DESCRIPTION:
XS GIS Cut Line= 3
       1551232.6      1093984.67      1550811.34      1093979.27
      1550398.19      1093990.08
#Sta/Elev= 30
  4576.8  833.96  4718.4  831.76  4766.1  832.114767.326 829.1354797.576 825.832
4850.913 824.1034865.506 822.8354904.031 814.1534909.492 813.6414920.245 810.455
4934.445 808.8964952.569 803.262  4974.5 798.0444980.428 795.9745008.932 794.421
  5016.3 793.2775021.068 793.6625022.041 795.413  5025.5 797.9675030.013 800.206
5031.502 812.5465052.072 813.1335074.556 811.0115079.796 818.8435101.183  832.15
 5112.93 837.7035124.261  838.18  5233.5  836.85  5291.6   844.5  5411.4  853.03
#Mann= 3 ,-1,0
  4576.8     .11       0  4974.5     .04       0  5025.5      .1       0
#XS Ineff= 2 , 0
       0    4850  833.26    5150       0  837.09
Permanent Ineff=
       F       F
Bank Sta=4974.5,5025.5
XS Rating Curve= 0 ,0
Exp/Cntr=0.5,0.3

--- GeorgesCreek.g03 (geometry) ---

Geom Title=Temporary Condition
Program Version=6.10

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
River Reach=Georges Creek   ,Reach-1

Type RM Length L Ch R = 1 ,7000    ,589,589,589
BEGIN DESCRIPTION:
Georges Creek 14.0
END DESCRIPTION:
XS GIS Cut Line= 3
        1550589.      1095675.48      1550326.46      1095246.59
      1550094.58      1095038.68
#Sta/Elev= 17
  4556.7  822.41  4605.2  816.38  4628.3  816.08  4700.4  811.87  4833.5  808.13
  4919.6  811.65  4979.3  800.26  4981.3  796.26  5018.7  796.26  5020.7  800.26
  5026.3  805.58    5040  811.19  5055.6  811.77  5088.2  812.32  5107.6  812.04
  5151.9  820.68    5260     821
#Mann= 3 ,-1,0
  4556.7     .15       0  4979.3    .042       0  5020.7     .11       0
Bank Sta=4979.3,5020.7
XS Rating Curve= 0 ,0
Exp/Cntr=0.5,0.3

Type RM Length L Ch R = 1 ,6420    ,39,39,39
BEGIN DESCRIPTION:
Georges Creek 13.0
END DESCRIPTION:
XS GIS Cut Line= 2
    1551220.9265    1095051.0574    1550283.4392    1094621.2055
#Sta/Elev= 30
  4371.5  820.81  4433.8  814.98  4495.2  811.66  4533.4  810.26  4616.9  809.07
  4632.3  808.36  4636.2  809.08  4704.6  808.97  4834.8  810.23  4898.1  808.37
  4934.9  807.95  4956.2  808.43    4960 804.386  4964.6  799.49  4966.7  796.35
  4979.9  796.17  4995.6  796.81  5002.7  799.36  5005.4  802.75  5011.2  803.51
  5029.2  802.86  5043.6  811.39  5054.6   819.6  5103.7  820.42  5126.7  820.95
  5183.9  823.12  5310.8  829.46  5363.2  836.01  5391.2  837.76  5402.8  837.94
#Mann= 3 ,-1,0
  4371.5     .15       0  4956.2    .042       0  5103.7      .1       0
#XS Ineff= 2 , 0
       0 4841.47  821.36 5187.47       0  825.06
Permanent Ineff=
       F       F
Bank Sta=4960,5005.4
XS Rating Curve= 0 ,0
Exp/Cntr=0.5,0.3

Type RM Length L Ch R = 1 ,6381    ,86,86,86
BEGIN DESCRIPTION:
Georges Creek 13.0
END DESCRIPTION:
XS GIS Cut Line= 4
    1551237.1813    1095015.6063    1551237.1813    1095015.6063
1550554.584369411094702.62543343     1550299.694    1094585.7544
#Sta/Elev= 30
 4371.75  828.13 4444.85  824.65 4534.65  821.27 4634.78     819  4738.6  819.23
 4840.41  820.05  4923.9  819.71 4943.91  817.68 4960.24  806.93 4962.95  805.66
 4977.47   805.5 4982.89  800.77 4990.11  797.98 4996.65  797.92 5009.56  795.99
 5013.89  795.89 5029.15  796.95 5038.42  804.34 5042.18  805.83 5053.51  811.72
 5061.54  813.47 5065.82  813.87 5075.89  817.65 5087.13  821.11 5093.13   821.9
  5099.6  821.56 5139.15  822.93 5258.34  828.34 5271.38  828.17 5403.09  834.67
#Mann= 3 ,-1,0
 4371.75     .15       0 4977.47    .042       0 5038.42      .1       0
#XS Ineff= 2 , 0
     .25 4898.55  824.38 5072.55     .25  824.38
Permanent Ineff=
       F       F
Bank Sta=4977.47,5038.42
XS Rating Curve= 0 ,0
Exp/Cntr=0.5,0.3

Type RM Length L Ch R = 3 ,6315    ,,,
BEGIN DESCRIPTION:
Old Easley Hwy. - TOR
Structure ID: LDS_GC_04
Approximate Survey Structure
END DESCRIPTION:
Bridge Culvert--1,0,-1,-1, 0
Deck Dist Width WeirC Skew NumUp NumDn MinLoCord MaxHiCord MaxSubmerge Is_Ogee
38,36,3,0, 101, 101, , , , 0, 1,1,,
  4371.5 4378.964382.864  4383.24388.4614401.3384406.5864410.5254412.3794421.558
4430.0454437.1174437.8764438.4174447.9654448.7614453.8394462.2044470.3554475.687
4482.0684486.5414487.4414489.5424495.8114503.5574510.1144521.8094532.3244537.422
4540.8064541.3474550.2264559.6414591.9224605.2024617.6154633.6334644.0624644.813
 4655.424664.4944709.4794742.1454746.127 4751.74 4778.774798.7544815.0954839.658
4843.5694843.5874844.2284855.3414866.5874892.0544910.732  4922.8  4922.8 4937.47
4939.7364942.1074944.6184944.618  5077.3  5077.3 5091.47 5091.475100.2975100.725
5106.5755133.0045147.8345158.4895186.0875192.0735192.2155192.2615192.3645192.501
5192.5495192.7075210.937  5213.15239.255 5262.155281.9165292.364 5292.425292.582
5298.8485318.9895350.7345367.0135391.2875397.3595399.5415401.6355406.1855419.167
5434.951
 828.775 828.501 828.358 828.346 828.163 827.713 827.529 827.391 827.326 827.003
 826.705 826.455 826.428 826.407 826.071 826.042  825.86 825.561 825.269 825.078
 824.849 824.689 824.657 824.606 824.453 824.265 824.105  823.82 823.563 823.439
 823.359 823.346 823.186 823.017 822.436 822.197 821.973 821.683 821.491  821.49
 821.475 821.463 821.402 821.358 821.343 821.382 821.572 821.712 821.827 821.999
 822.027 822.027 822.029 822.062 822.095  822.17 822.225  822.28  822.28  822.29
  822.31 822.317 822.326 822.326  822.33  822.33  822.34  822.34 822.369 822.373
 822.554 823.372 823.831 824.161 825.016 825.201 825.206 825.208 825.212 825.219
 825.221 825.229 826.136 826.244 827.542 828.678 829.659 830.178 830.178 830.188
 830.506 831.526 833.135  833.96  835.19 835.498 835.609 835.714 835.941 836.588
 837.375
                                                                                
                                                                                
                                                                                
                                                                                
                                                                                
                                                           820.2   820.2  820.21
  820.23  820.24  820.25  820.25  820.25  820.25  820.26
                                                                                
                                                                                
                                                                                
        
  4371.5 4378.964382.864  4383.24388.4614401.3384406.5864410.5254412.3794421.558
4430.0454437.1174437.8764438.4174447.9654448.7614453.8394462.2044470.3554475.687
4482.0684486.5414487.4414489.5424495.8114503.5574510.1144521.8094532.3244537.422
4540.8064541.3474550.2264559.6414591.9224605.2024617.6154633.6334644.0624644.813
 4655.424664.4944709.4794742.1454746.127 4751.74 4778.774798.7544815.0954839.658
4843.5694843.5874844.2284855.3414866.5874892.0544910.732  4922.8  4922.8 4937.47
4939.7364942.1074944.6184944.618  5077.3  5077.3 5091.47 5091.475100.2975100.725
5106.5755133.0045147.8345158.4895186.0875192.0735192.2155192.2615192.3645192.501
5192.5495192.7075210.937  5213.15239.255 5262.155281.9165292.364 5292.425292.582
5298.8485318.9895350.7345367.0135391.2875397.3595399.5415401.6355406.1855419.167
5434.951
 828.775 828.501 828.358 828.346 828.163 827.713 827.529 827.391 827.326 827.003
 826.705 826.455 826.428 826.407 826.071 826.042  825.86 825.561 825.269 825.078
 824.849 824.689 824.657 824.606 824.453 824.265 824.105  823.82 823.563 823.439
 823.359 823.346 823.186 823.017 822.436 822.197 821.973 821.683 821.491  821.49
 821.475 821.463 821.402 821.358 821.343 821.382 821.572 821.712 821.827 821.999
 822.027 822.027 822.029 822.062 822.095  822.17 822.225  822.28  822.28  822.29
  822.31 822.317 822.326 822.326  822.33  822.33  822.34  822.34 822.369 822.373
 822.554 823.372 823.831 824.161 825.016 825.201 825.206 825.208 825.212 825.219
 825.221 825.229 826.136 826.244 827.542 828.678 829.659 830.178 830.178 830.188
 830.506 831.526 833.135  833.96  835.19 835.498 835.609 835.714 835.941 836.588
 837.375
                                                                                
                                                                                
                                                                                
                                                                                
                                                                                
                                                           820.2   820.2  820.21
  820.23  820.24  820.25  820.25  820.25  820.25  820.26
                                                                                
                                                                                
                                                                                
        
Pier Skew, UpSta & Num, DnSta & Num=  ,4944.8, 2 ,4944.8, 2 , 0 , 0 , 0 ,0,0
    1.75    1.75
  809.22   820.8
    1.75    1.75
  805.66   820.8
Pier Skew, UpSta & Num, DnSta & Num=  ,4966.8, 2 ,4966.8, 2 , 0 , 0 , 0 ,0,0
    1.75    1.75
  810.17   820.8
    1.75    1.75
  805.03   820.8
Pier Skew, UpSta & Num, DnSta & Num=  ,4988.8, 2 ,4988.8, 2 , 0 , 0 , 0 ,0,0
    1.75    1.75
   794.5   820.8
    1.75    1.75
  794.25   820.8
Pier Skew, UpSta & Num, DnSta & Num=  ,5010.8, 2 ,5010.8, 2 , 0 , 0 , 0 ,0,0
    1.75    1.75
   794.5   820.8
    1.75    1.75
  794.25   820.8
Pier Skew, UpSta & Num, DnSta & Num=  ,5032.8, 2 ,5032.8, 2 , 0 , 0 , 0 ,0,0
    1.75    1.75
   811.8   820.8
    1.75    1.75
  803.26   820.8
Pier Skew, UpSta & Num, DnSta & Num=  ,5054.8, 2 ,5054.8, 2 , 0 , 0 , 0 ,0,0
    1.75    1.75
  818.59   820.8
    1.75    1.75
  815.79   820.8
Abutment Skew #Up #Dn= , 2 , 2
  4922.8 4943.37
     820     808
  4922.8 4943.37
     820     808
Abutment Skew #Up #Dn= , 2 , 2
 5090.47 5091.47
  819.22  820.08
  5076.3  5077.3
  819.22  820.08
BR Coef=-1 ,-1 , 0 ,1.25, 0 ,,,0.8,0,2,0,
WSPro=,,,, 1 ,,,, 0 ,,,, 0 ,,,,-1 ,-1 ,-1 , 0 , 0 , 0 , 0 , 0
BC Design=,, 0 ,, 0 ,,,,,,
BC HTab HWMax=843.14
BC Use User HTab Curves=0
BC User HTab FreeFlow(D)= 0

Type RM Length L Ch R = 1 ,6220    ,260,260,260
XS GIS Cut Line= 2
    1551320.6064    1094872.9437    1550360.5379    1094437.7468
#Sta/Elev= 30
    4430     845    4665  844.67 4690.89  843.94 4699.84  836.89 4710.87  834.46
 4742.87   814.6 4748.83  811.77 4758.32  809.73  4785.9  808.23 4811.28  809.69
 4959.12  810.55 4963.54  809.08 4967.95  803.04 4975.67  801.63 4983.62  798.23
 5010.98  797.48  5015.4  798.64 5018.98  801.76 5022.02  806.74    5025   809.4
 5036.29  811.13  5050.7  822.32 5069.46  833.99 5078.43  832.24 5159.93  833.15
 5200.76   835.3 5242.48  839.45 5285.72  839.07 5311.09  843.73  5337.7   846.4
#Mann= 4 ,-1,0
    4430     .15       0    4665     .15       0 4975.67    .045       0
 5018.98     .12       0
#XS Ineff= 2 , 0
       0  4774.8  820.36  5225.3       0  820.36
Permanent Ineff=
       F       F
Bank Sta=4975.67,5018.98
XS Rating Curve= 0 ,0
Exp/Cntr(USF)=0,0
Exp/Cntr=0.5,0.3

Type RM Length L Ch R = 1 ,5960    ,57.6,57.6,57.6
BEGIN DESCRIPTION:
Georges Creek 12.0
END DESCRIPTION:
XS GIS Cut Line= 4
      1551040.87      1094403.23      1550762.74      1094346.52
      1550552.11      1094357.321550540.936689951094357.89290865
#Sta/Elev= 27
  4710.1  823.37  4759.9  810.24  4764.7  810.474842.529 809.2544892.841 808.599
4932.809 808.6794944.874 808.8964977.175 808.5334988.165 800.3794989.785 798.446
4990.566  796.734992.082 796.7645008.815 796.2845017.452 796.7655027.048 797.088
 5029.24 799.4165038.279 809.0145040.111 810.6495045.509 814.2795067.002  827.08
5071.343 830.384 5074.81 832.1195082.657 836.561 5087.96 835.7115117.904 836.397
5133.088  836.87    5210   836.9
#Mann= 3 ,-1,0
  4710.1     .15       04988.165     .04       0 5029.24     .12       0
Bank Sta=4988.165,5029.24
XS Rating Curve= 0 ,0
Exp/Cntr=0.5,0.3

Type RM Length L Ch R = 1 ,5902    ,102,102,102
XS GIS Cut Line= 2
1551186.417496921094302.36684743 1550486.40119381094275.80076382
#Sta/Elev= 30
       0  831.05   11.93  826.55   57.96  815.87   64.96  813.42   78.97  814.07
   90.98  812.94   258.1  809.35  298.13  809.59  326.15  808.09   389.3  808.28
  400.21  804.42  404.21  800.83  407.21  798.55  411.21  797.05   416.3  796.76
  431.23  798.97  435.89  797.44  443.24  797.32  448.24  800.99  452.24  804.99
  459.25  809.68  472.22  810.58  484.27   814.3  501.28  824.87  512.29  833.81
  519.29  836.53  542.31  835.31  624.37  840.46   675.4  840.35  700.52  842.41
#Mann= 3 ,-1,0
       0     .15       0  404.21    .045       0  448.24     .12       0
Bank Sta=404.21,448.24
XS Rating Curve= 0 ,0
Exp/Cntr(USF)=0,0
Exp/Cntr=0.3,0.1

Type RM Length L Ch R = 1 ,5800    ,42,42,42
BEGIN DESCRIPTION:
Georges Creek 11.5
END DESCRIPTION:
XS GIS Cut Line= 2
      1551170.49       1094192.6    1550419.6349    1094182.1911
#Sta/Elev= 30
    4603  825.18    4603  825.16  4608.2  822.06    4613  820.71  4657.6  817.26
    4683  818.22  4708.6  814.43  4780.6  811.83  4792.1  811.52  4832.7  812.66
  4907.8  808.45  4966.9  807.99  4974.5  803.83  4982.9  797.01    4993  797.36
  5001.3   796.6  5016.6  796.52  5023.5  797.02  5031.6   804.9  5035.6  809.22
  5083.5  811.55  5090.9  813.53  5101.4  812.92  5126.7  830.04  5144.9  837.21
  5273.9  840.19  5282.4  841.34  5339.4  844.16  5348.8  845.35  5353.9  848.08
#Mann= 3 ,-1,0
    4603     .13       0  4974.5     .04       0  5031.6      .1       0
#XS Ineff= 2 , 0
       0    4816  834.26    5184       0   837.8
Permanent Ineff=
       F       F
Bank Sta=4974.5,5031.6
XS Rating Curve= 0 ,0
Exp/Cntr=0.5,0.3

Type RM Length L Ch R = 1 ,5758    ,127,127,127
BEGIN DESCRIPTION:
Georges Creek 11.5
END DESCRIPTION:
XS GIS Cut Line= 2
    1551171.0722     1094150.604     1550420.217    1094140.1951
#Sta/Elev= 30
    4603  832.37 4606.91  832.37 4618.43  826.94 4630.42  825.06 4681.53  823.56
 4701.16  820.84 4730.48  819.92 4766.87  823.82 4790.84  823.76 4868.79  820.39
 4881.33  818.91 4894.71  814.58 4906.78  808.31 4968.19  807.45  4974.5  803.62
 4985.11  796.37 5006.02  796.03 5020.42   796.4  5031.6  805.75  5038.1     810
  5053.6  812.12 5086.16  821.84 5136.57  823.65 5159.13  830.65 5165.88  835.65
 5179.53  837.91 5227.28  837.57 5240.96  838.66 5271.01  844.59 5353.93  848.93
#Mann= 3 ,-1,0
    4603     .13       0  4974.5     .04       0  5031.6      .1       0
#XS Ineff= 2 , 0
       0 4895.27  834.26    5101       0  834.26
Permanent Ineff=
       F       F
Bank Sta=4974.5,5031.6
XS Rating Curve= 0 ,0
Exp/Cntr=0.5,0.3

Type RM Length L Ch R = 3 ,5677    ,,,
BEGIN DESCRIPTION:
US Hwy 123 (Georges Cr.) - TOR
Structure ID: LDS_GC_03
Approximate Survey Structure
END DESCRIPTION:
Bridge Culvert--1,0,-1,-1, 0
Deck Dist Width WeirC Skew NumUp NumDn MinLoCord MaxHiCord MaxSubmerge Is_Ogee
1,125,3,0, 20, 20, , , , 0, 1,1,,
    4603 4630.26 4630.73 4680.33 4730.12 4780.09  4830.3  4883.7    4900    4900
    5100    5100 5146.87 5196.91 5246.78 5246.78 5297.07 5297.07 5346.71 5396.73
 839.271 838.263 838.248 836.737 835.487 834.602 834.282 834.257 834.257 834.257
 837.904 837.904 839.803 842.112 844.467 844.467 846.856 846.856 849.443 851.924
                                                                           831.5
  835.14
    4603 4630.26 4630.73 4680.33 4730.12 4780.09  4830.3  4883.7    4900    4900
    5100    5100 5146.87 5196.91 5246.78 5246.78 5297.07 5297.07 5346.71 5396.73
 839.271 838.263 838.248 836.737 835.487 834.602 834.282 834.257 834.257 834.257
 837.904 837.904 839.803 842.112 844.467 844.467 846.856 846.856 849.443 851.924
                                                                           831.5
  835.14
Pier Skew, UpSta & Num, DnSta & Num=  ,4925, 2 ,4925, 2 , 0 , 0 , 0 ,0,0
    2.33    2.33
  808.63     832
    2.33    2.33
  810.79     832
Pier Skew, UpSta & Num, DnSta & Num=  ,4962, 2 ,4962, 2 , 0 , 0 , 0 ,,
       5       5
     800     833
       5       5
     800     833
Pier Skew, UpSta & Num, DnSta & Num=  ,4975, 2 ,4975, 2 , 0 , 0 , 0 ,0,0
    2.33    2.33
  805.77     833
    2.33    2.33
  805.52     833
Pier Skew, UpSta & Num, DnSta & Num=  ,5025, 2 ,5025, 2 , 0 , 0 , 0 ,0,0
    2.33    2.33
  805.77   834.6
    2.33    2.33
  805.52   834.6
Pier Skew, UpSta & Num, DnSta & Num=  ,5067, 2 ,5067, 2 , 0 , 0 , 0 ,,
       5       5
     800     835
       5       5
     800     835
Pier Skew, UpSta & Num, DnSta & Num=  ,5075, 2 ,5075, 2 , 0 , 0 , 0 ,0,0
    2.33    2.33
  809.44   835.6
    2.33    2.33
  815.52   835.6
Abutment Skew #Up #Dn= , 10 , 10
    4900 4902.39 4904.05 4907.63 4908.73 4911.98 4923.34 4925.11 4929.03 4941.87
 830.465 830.465  827.77 826.686 826.475 824.555 817.377  816.54 814.314 808.123
    4900 4902.39 4904.05 4907.63 4908.73 4911.98 4923.34 4925.11 4929.03 4941.87
 830.465 830.465  827.77 826.686 826.475 824.555 817.377  816.54 814.314 808.123
Abutment Skew #Up #Dn= , 8 , 8
    5054 5054.43 5060.64 5063.99 5072.63 5074.05 5075.51    5100
     810  811.08   816.1  818.38  823.04  823.92  824.56  833.04
    5054 5054.43 5060.64 5063.99 5072.63 5074.05 5075.51    5100
     810  811.08   816.1  818.38  823.04  823.92  824.56  833.04
BR Coef=-1 ,-1 , 0 ,1.25, 0 ,,,0.8,0,2,0,
WSPro=,,,, 1 ,,,, 0 ,,,, 0 ,,,,-1 ,-1 ,-1 , 0 , 0 , 0 , 0 , 0
BC Design=,, 0 ,, 0 ,,,,,,
BC HTab HWMax=845.29
BC Use User HTab Curves=0
BC User HTab FreeFlow(D)= 0

Type RM Length L Ch R = 1 ,5631    ,43,43,43
BEGIN DESCRIPTION:
Georges Creek 11.5
END DESCRIPTION:
XS GIS Cut Line= 2
    1551172.8326    1094023.6162    1550421.9774    1094013.2073
#Sta/Elev= 30
    4628  836.91 4654.91  835.79  4704.8  834.99 4752.48  834.99  4762.8  834.47
 4768.53  832.21 4804.86  830.19 4896.89  829.58 4911.73  826.97 4931.69  814.73
 4946.53  808.17 4956.48   805.8 4971.03  806.29 4979.42  799.29 4982.84  796.23
 5003.29  795.28  5021.2  796.46 5021.99  797.91 5024.45  799.92 5034.19  808.03
 5065.63  814.83 5102.32  833.27  5110.2  835.63 5306.74  846.23 5315.57  845.47
 5327.31  847.28 5339.32  848.04 5365.62  849.05 5372.73  848.45 5378.93  848.88
#Mann= 3 ,-1,0
    4628     .13       0 4979.42     .04       0 5024.45      .1       0
#XS Ineff= 2 , 0
       0    4891   831.5    5123       0   831.5
Permanent Ineff=
       F       F
Bank Sta=4979.42,5024.45
XS Rating Curve= 0 ,0
Exp/Cntr=0.5,0.3

Type RM Length L Ch R = 1 ,5588    ,588,588,588
BEGIN DESCRIPTION:
Georges Creek 11.0
END DESCRIPTION:
XS GIS Cut Line= 3
       1551232.6      1093984.67      1550811.34      1093979.27
      1550398.19      1093990.08
#Sta/Elev= 30
  4576.8  833.96  4718.4  831.76  4766.1  832.114767.326 829.1354797.576 825.832
4850.913 824.1034865.506 822.8354904.031 814.1534909.492 813.6414920.245 810.455
4934.445 808.8964952.569 803.262  4974.5 798.0444980.428 795.9745008.932 794.421
  5016.3 793.2775021.068 793.6625022.041 795.413  5025.5 797.9675030.013 800.206
5031.502 812.5465052.072 813.1335074.556 811.0115079.796 818.8435101.183  832.15
 5112.93 837.7035124.261  838.18  5233.5  836.85  5291.6   844.5  5411.4  853.03
#Mann= 3 ,-1,0
  4576.8     .11       0  4974.5     .04       0  5025.5      .1       0
#XS Ineff= 2 , 0
       0    4850  833.26    5150       0  837.09
Permanent Ineff=
       F       F
Bank Sta=4974.5,5025.5
XS Rating Curve= 0 ,0
Exp/Cntr=0.5,0.3

--- GeorgesCreek.g09 (geometry) ---

Geom Title=Unrestricted
Program Version=6.10

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
River Reach=Georges Creek   ,Reach-1

Type RM Length L Ch R = 1 ,58431   ,83,83,83
BEGIN DESCRIPTION:
Georges Creek 117.5
END DESCRIPTION:
XS GIS Cut Line= 3
      1515124.85      1098241.73      1515027.31      1098179.35
      1514939.98      1098114.71
#Sta/Elev= 10
  4884.9 1016.51  4972.6 1006.94  4998.2  999.52    4999  998.02    5001  998.02
  5001.8  999.52  5031.8 1004.46  5045.6 1007.33    5059 1008.37  5109.4 1023.85
#Mann= 3 ,-1,0
  4884.9     .15       0  4998.2     .05       0  5001.8     .15       0
Bank Sta=4998.2,5001.8
XS Rating Curve= 0 ,0
Exp/Cntr=0.3,0.1

Type RM Length L Ch R = 1 ,58348   ,81,81,81
BEGIN DESCRIPTION:
Georges Creek 117
END DESCRIPTION:
XS GIS Cut Line= 3
       1515149.8      1098152.13      1515064.74      1098105.63
      1514991.02      1098068.21
#Sta/Elev= 10
  4909.2 1016.78  4937.1 1012.75  4974.5 1004.81    4990 1000.12  4997.5  998.52
  5002.5  998.52    5010 1000.12  5048.5 1006.44  5049.5 1006.61  5088.8 1021.44
#Mann= 3 ,-1,0
  4909.2     .15       0    4990     .05       0    5010     .15       0
#XS Ineff= 2 , 0
Permanent Ineff=
       F       F
Bank Sta=4990,5010
XS Rating Curve= 0 ,0
Exp/Cntr=0.3,0.1

Type RM Length L Ch R = 1 ,58267   ,270,270,270
BEGIN DESCRIPTION:
Georges Creek 116.5
END DESCRIPTION:
XS GIS Cut Line= 3
      1515221.26      1098102.23      1515107.84      1098037.58
      1515018.24      1098001.29
#Sta/Elev= 14
  4853.8 1016.58    4862 1016.08    4917 1013.86  4922.6 1013.28  4927.5 1012.19
  4960.5 1004.33  4984.4 1001.17    4990 1000.02  4997.5  998.42  5002.5  998.42
    5010 1000.02  5035.7 1004.77  5058.6  1015.9    5081 1025.42
#Mann= 3 ,-1,0
  4853.8     .15       0    4990     .05       0    5010     .15       0
#XS Ineff= 2 , 0
Permanent Ineff=
       F       F
Bank Sta=4990,5010
XS Rating Curve= 0 ,0
Exp/Cntr=0.3,0.1

Type RM Length L Ch R = 1 ,57997   ,535,535,535
BEGIN DESCRIPTION:
Georges Creek 116.0
END DESCRIPTION:
XS GIS Cut Line= 3
        1515425.        1098025.      1515288.85      1097858.76
      1515176.88      1097746.14
#Sta/Elev= 16
  4785.1 1019.58  4797.4 1019.44  4884.1 1009.53  4947.1 1004.23  4948.5 1003.97
  4998.5  992.85  4999.2  991.35  5000.8  991.35  5001.5  992.85    5009  992.85
  5030.6  995.03  5043.8  997.34  5060.1  999.56  5099.6 1008.74  5128.3 1018.37
  5158.8 1023.97
#Mann= 3 ,-1,0
  4785.1     .15       0  4998.5     .05       0  5001.5     .15       0
Bank Sta=4998.5,5001.5
XS Rating Curve= 0 ,0
Exp/Cntr=0.3,0.1

Type RM Length L Ch R = 1 ,57462   ,103,103,103
BEGIN DESCRIPTION:
Georges Creek 115.0
END DESCRIPTION:
XS GIS Cut Line= 3
      1515744.85      1097801.92       1515691.6      1097571.18
      1515580.04       1097251.7
#Sta/Elev= 19
  4754.5 1013.82  4767.3 1013.05  4794.1 1009.98    4811 1009.32  4813.6 1009.34
  4958.5  996.44  4990.1  994.11  4997.3  988.91  5002.8  988.91  5009.9  994.11
  5037.8  996.35  5043.2  997.88  5046.2  998.53  5053.5  998.97    5072 1000.55
  5092.3 1003.09  5138.4 1007.37  5251.7 1020.81  5329.7 1026.57
#Mann= 3 ,-1,0
  4754.5     .15       0  4990.1     .05       0  5009.9     .15       0
#XS Ineff= 2 , 0
Permanent Ineff=
       F       F
Bank Sta=4990.1,5009.9
XS Rating Curve= 0 ,0
Exp/Cntr=0.3,0.1

Type RM Length L Ch R = 1 ,57359   ,362,362,362
BEGIN DESCRIPTION:
Georges Creek 114.5
END DESCRIPTION:
XS GIS Cut Line= 3
      1515869.09       1097779.1      1515787.95      1097545.83
      1515671.32      1097239.02
#Sta/Elev= 27
  4750.1 1013.49  4765.2  1009.8  4785.2 1007.57  4812.1 1006.77  4814.9 1006.52
    4837 1007.39  4903.4  998.21  4919.2  997.23  4952.6  996.33  4965.9   996.7
  4975.9  993.29    4991  993.85  4997.5  988.65  5002.5  988.65    5009  993.85
  5020.2  991.61  5026.4  993.89  5030.1  994.06  5076.3 1001.85  5107.5 1007.88
  5127.2 1010.52  5150.2 1012.39  5160.1 1014.14  5190.4 1014.43  5273.4 1024.49
  5314.6 1028.58  5325.3 1029.29
#Mann= 3 ,-1,0
  4750.1     .14       0    4991     .05       0    5009     .14       0
#XS Ineff= 2 , 0
Permanent Ineff=
       F       F
Bank Sta=4991,5009
XS Rating Curve= 0 ,0
Exp/Cntr=0.3,0.1

Type RM Length L Ch R = 1 ,56997   ,450,450,450
BEGIN DESCRIPTION:
Georges Creek 114.0
END DESCRIPTION:
XS GIS Cut Line= 3
      1516059.26       1097850.1      1516138.96       1097478.3
      1516097.29      1097264.38
#Sta/Elev= 22
  4619.8  1012.3  4621.7 1012.14  4655.2 1010.44  4675.9 1009.86  4701.3 1010.01
  4757.4 1005.27  4802.4 1004.88  4834.9  1001.4  4855.7 1000.08  4934.4   992.8
  4949.9  991.81  4977.8  987.81  4997.3  983.81  4998.6  982.31  5001.4  982.31
  5002.7  983.81  5025.3  988.55  5039.4  991.14  5057.2  993.16  5140.1 1007.72
  5181.6 1012.19  5217.9 1018.27
#Mann= 3 ,-1,0
  4619.8     .15       0  4997.3     .05       0  5002.7     .15       0
Bank Sta=4997.3,5002.7
XS Rating Curve= 0 ,0
Exp/Cntr=0.3,0.1

Type RM Length L Ch R = 1 ,56547   ,143,143,143
BEGIN DESCRIPTION:
Georges Creek 113.0
END DESCRIPTION:
XS GIS Cut Line= 4
       1516404.1      1097591.47      1516556.52      1097397.78
      1516619.62      1097241.56       1516553.7      1097180.71
#Sta/Elev= 30
  4716.9  997.96  4723.5  997.52  4756.4  994.47  4780.4  993.44  4786.9  993.37
  4790.1  992.88  4797.7  993.07  4799.4  992.97  4810.9  991.78  4815.2  991.62
  4830.9  990.37  4838.1  990.16  4852.9  989.15  4856.4   989.1  4917.1  986.99
  4928.6     986    4951  984.67  4963.3  983.68  4992.8  983.83    4997  980.53
    5003  980.53  5007.2  983.83    5033  984.42    5048  988.66  5095.4  991.65
  5131.8   993.1  5132.1  993.11  5158.3  996.38  5219.8 1002.43  5221.6 1002.56
#Mann= 3 ,-1,0
  4716.9     .15       0  4992.8     .05       0  5007.2     .15       0
#XS Ineff= 2 , 0
Permanent Ineff=
       F       F
Bank Sta=4992.8,5007.2
XS Rating Curve= 0 ,0
Exp/Cntr=0.3,0.1

Type RM Length L Ch R = 1 ,56404   ,548,548,548
BEGIN DESCRIPTION:
Georges Creek 112.5
END DESCRIPTION:
XS GIS Cut Line= 4
      1516544.98      1097602.71      1516675.84      1097358.83
      1516669.38      1097320.07      1516891.25      1096947.79
#Sta/Elev= 30
  4700.5  996.58  4789.8  992.98  4794.9  992.65  4818.3  991.91  4819.1  991.97
  4822.2  991.72  4849.6  988.46  4925.4  986.77  4933.2  986.79  4938.9  985.76
  4977.2  986.08  4992.5  980.63  4996.5  979.13    5004  979.13  5007.5  980.63
  5010.6  980.87  5016.5  982.73  5032.7  982.71  5068.8  986.12  5078.4  986.03
    5088  986.71  5197.9  989.63  5210.1  990.27  5218.2   990.9  5323.2  991.14
  5343.5  990.15  5370.8  989.71  5382.3  990.39    5408  991.11  5449.9  990.67
#Mann= 3 ,-1,0
  4700.5     .15       0  4992.5     .05       0  5007.5     .15       0
#XS Ineff= 2 , 0
Permanent Ineff=
       F       F
Bank Sta=4992.5,5007.5
XS Rating Curve= 0 ,0
Exp/Cntr=0.3,0.1

Type RM Length L Ch R = 1 ,55856   ,130,130,130
BEGIN DESCRIPTION:
Georges Creek 112.0
END DESCRIPTION:
XS GIS Cut Line= 4
      1517281.41      1097454.55      1517278.87       1097216.2
      1517177.45      1097086.89      1516863.04      1096757.26
#Sta/Elev= 30
  4600.2 1003.02  4611.1    1003  4620.7  999.63    4622  999.59  4678.2  995.06
  4702.9  993.77  4720.3   991.4  4742.2   990.4  4746.4  989.41  4787.7  986.64
  4801.4  986.24  4838.6  986.26  4973.1  984.71    4983   981.9  4995.5   976.4
  5004.5   976.4    5017   981.9  5027.3  983.08  5036.4  983.36  5312.2  985.64
  5332.1  985.93  5345.5  986.48  5369.9  990.07  5384.5  990.45  5387.9   990.4
    5398  991.93  5419.9  994.79  5430.8  995.43  5441.9  994.64  5458.5  994.86
#Mann= 3 ,-1,0
  4600.2     .15       0    4983     .05       0    5017     .15       0
#XS Ineff= 2 , 0
Permanent Ineff=
       F       F
Bank Sta=4983,5017
XS Rating Curve= 0 ,0
Exp/Cntr=0.3,0.1

Type RM Length L Ch R = 1 ,55726   ,278,278,278
BEGIN DESCRIPTION:
Georges Creek 111.5
END DESCRIPTION:
XS GIS Cut Line= 3
      1517377.76       1097436.8      1517400.58       1097173.1
      1516999.96       1096716.7
#Sta/Elev= 28
  4590.6  991.83  4640.5   988.9  4641.8  988.77  4644.4  988.79  4712.4  986.32
    4754  986.62  4767.1  986.18  4791.3   984.5    4801  985.57  4838.3  978.32
  4855.3  979.09  4930.1  980.25    4983  979.58  4995.5  976.08  5004.5  976.08
    5017  979.58  5048.8  977.63  5083.3  976.56  5088.7  976.79  5099.1  976.82
  5131.4  976.15  5173.8  977.98  5187.6  976.93  5273.2  979.99  5283.6  980.64
    5299  982.08    5319  983.32    5432  987.19
#Mann= 3 ,-1,0
  4590.6     .15       0    4983     .05       0    5017     .15       0
#XS Ineff= 2 , 0
Permanent Ineff=
       F       F
Bank Sta=4983,5017
XS Rating Curve= 0 ,0
Exp/Cntr=0.3,0.1

Type RM Length L Ch R = 1 ,55448   ,76,76,76
BEGIN DESCRIPTION:
Georges Creek 111.0
END DESCRIPTION:
XS GIS Cut Line= 3
      1517289.01      1097576.26      1517534.97      1097213.67
      1517633.85      1097041.25
#Sta/Elev= 30
  4566.1 1009.04  4605.3 1006.92  4612.1 1006.21  4637.1 1002.13  4659.7  999.14
  4678.9  996.13  4704.4  993.38    4717  992.63  4745.5  991.65    4769  988.63
  4787.6  987.64  4805.6   987.4  4811.9  987.46  4831.1  987.27  4840.2  986.96
  4888.2  986.32  4898.8  984.67    4924  981.51  4934.5   981.3  4949.6  981.69
    4992   981.5    4998   974.4    5002   974.4    5008   981.5  5044.6  990.13
  5046.1  990.31  5109.9  995.48  5169.1 1006.94  5200.5 1008.17    5203 1008.33
#Mann= 3 ,-1,0
  4566.1     .15       0    4992     .05       0    5008     .15       0
#XS Ineff= 2 , 0
Permanent Ineff=
       F       F
Bank Sta=4992,5008
XS Rating Curve= 0 ,0
Exp/Cntr=0.3,0.1

Type RM Length L Ch R = 1 ,55372   ,179,179,179
BEGIN DESCRIPTION:
Georges Creek 110.5
END DESCRIPTION:
XS GIS Cut Line= 4
       1517344.8      1097616.83      1517552.71      1097332.84
      1517674.42      1097122.39       1517687.1      1097056.46
#Sta/Elev= 30
    4560 1006.64  4595.1  1003.9  4626.7  999.36  4665.3  998.46  4675.9  996.62
  4684.5  996.35  4730.9  989.97  4774.3  989.87  4783.9  989.32  4788.5  988.57
  4808.7  987.81  4814.2  987.86  4827.4  986.86  4867.2  987.47  4896.7  981.74
  4916.8  979.86  4923.4   979.8    4948  978.39  4952.7  977.84    4992  978.03
    4998  970.93    5002  970.93    5008  978.03  5036.5  984.17  5067.3     994
    5090  994.93  5101.8  995.83  5167.9  998.12  5207.2 1008.21  5222.2 1009.62
#Mann= 3 ,-1,0
    4560     .15       0    4992     .05       0    5008     .15       0
#XS Ineff= 2 , 0
Permanent Ineff=
       F       F
Bank Sta=4992,5008
XS Rating Curve= 0 ,0
Exp/Cntr=0.3,0.1

Type RM Length L Ch R = 1 ,55193   ,164,164,164
BEGIN DESCRIPTION:
Georges Creek 110.0
END DESCRIPTION:
XS GIS Cut Line= 3
      1517536.27      1097928.13      1517787.49      1097241.47
       1517720.5      1097020.96
#Sta/Elev= 19
  4316.9  994.58  4321.2  994.35  4391.9  992.28  4576.3  990.44  4631.7  989.36
  4655.6  988.25  4816.2  983.16  4836.3  981.52  4858.9  980.38  4951.9  977.94
  4990.9   975.2  4994.8   969.9  5005.2   969.9  5009.1   975.2  5026.8  976.76
  5044.9  977.38  5048.1  977.26  5087.4  976.88  5201.9  990.07
#Mann= 3 ,-1,0
  4316.9    .145       0  4990.9    .049       0  5009.1    .145       0
#XS Ineff= 2 , 0
Permanent Ineff=
       F       F
Bank Sta=4990.9,5009.1
XS Rating Curve= 0 ,0
Exp/Cntr=0.3,0.1

Type RM Length L Ch R = 1 ,55029   ,532,532,532
BEGIN DESCRIPTION:
Georges Creek 109.5
END DESCRIPTION:
XS GIS Cut Line= 3
      1517644.46      1097990.65      1517923.68      1097348.14
      1518004.74      1096831.74
#Sta/Elev= 24
    4739  988.27  4798.4  981.92  4824.7  978.22  4931.2   976.8  4960.6  976.47
  4990.2  972.95  4994.4  969.65  5005.6  969.65  5009.8  972.95    5069  974.95
  5093.5  977.44  5104.3  976.97  5126.2  977.45  5154.8  980.74  5169.7  980.97
  5296.9   983.9  5352.3  982.95  5352.8  982.98  5358.1  983.35  5359.9  983.36
  5369.7  983.87  5372.3  983.84  5392.5  984.57  5419.6  982.15
#Mann= 3 ,-1,0
    4739     .14       0  4990.2    .048       0  5009.8     .14       0
#XS Ineff= 2 , 0
Permanent Ineff=
       F       F
Bank Sta=4990.2,5009.8
XS Rating Curve= 0 ,0
Exp/Cntr=0.3,0.1

Type RM Length L Ch R = 1 ,54497   ,320,320,320
BEGIN DESCRIPTION:
Georges Creek 109.0
END DESCRIPTION:
XS GIS Cut Line= 3
      1517616.27      1098342.77       1518347.8      1097604.42
      1518576.02      1097394.72
#Sta/Elev= 30
  3960.6 1007.51  3993.3 1004.04  4069.4  998.94  4122.7  997.42  4152.8  994.05
  4184.6  992.69  4228.3   989.6    4420  991.29  4558.2   985.8  4620.8  989.95
  4651.9  990.26  4667.6  991.39  4808.8   987.2  4816.4  986.71    4835  976.75
  4838.5  975.79  4912.1  974.54  4967.5  975.21  4996.1  966.08  4996.8  964.58
  5001.1  964.58  5002.1  966.08  5007.8  968.68  5021.3  971.88  5113.8  976.54
  5144.3  979.45  5190.6   985.2  5246.3  994.89  5266.1  995.63  5309.9  999.08
#Mann= 3 ,-1,0
  3960.6     .15       0  4996.1     .05       0  5002.1     .15       0
Bank Sta=4996.1,5002.1
XS Rating Curve= 0 ,0
Exp/Cntr=0.3,0.1

Type RM Length L Ch R = 1 ,54177   ,308,308,308
BEGIN DESCRIPTION:
Georges Creek 108.0
END DESCRIPTION:
XS GIS Cut Line= 4
      1518098.47      1098010.81      1518543.93      1097858.39
      1518625.26       1097778.4      1518571.28      1097560.32
#Sta/Elev= 30
  4472.8  990.51  4529.9  992.39  4553.4  991.87  4562.1  991.18  4582.8  991.62
  4640.1  989.13    4657  987.16  4697.9  980.98  4822.8  976.56  4873.4  976.61
  4918.3  975.31  4943.6  974.96  4961.4  973.71  4970.1  971.29  4979.6  967.71
    4985   967.9    4994     965    5006     965    5015   967.9  5032.8  971.72
  5051.1  971.22  5057.7  971.46  5071.7  973.17    5102  975.72  5131.8  976.66
  5150.8  976.23  5198.5  980.11  5213.3  982.85  5229.1  983.55  5282.4  987.41
#Mann= 3 ,-1,0
  4472.8     .15       0    4985     .05       0    5015     .15       0
#XS Ineff= 2 , 0
Permanent Ineff=
       F       F
Bank Sta=4985,5015
XS Rating Curve= 0 ,0
Exp/Cntr=0.3,0.1

Type RM Length L Ch R = 1 ,53869   ,211,211,211
BEGIN DESCRIPTION:
Georges Creek 107.9
END DESCRIPTION:
XS GIS Cut Line= 4
      1518506.19      1098494.64      1518840.58      1098043.69
      1518873.58      1097871.06       1518924.5      1097684.66
#Sta/Elev= 30
  4342.4  994.01    4370  993.67  4469.1  989.53  4515.5  986.03  4562.6  981.17
  4572.8  980.68  4679.9  979.58  4710.9  976.29  4775.3  975.91  4860.7   976.9
  4873.8  977.41  4901.2   975.3  4942.5  975.66  4960.3  975.12  4977.1  969.29
    4985  965.78    4994  961.88    5006  961.88    5015  965.78  5029.1  969.12
  5077.5  969.12  5094.2  973.92  5107.1  981.44  5138.6  981.63  5176.5  989.54
  5207.1  996.87  5225.9  998.88  5234.5  998.82  5259.3  1005.7  5272.8 1011.84
#Mann= 3 ,-1,0
  4342.4    .135       0    4985     .05       0    5015    .145       0
#XS Ineff= 2 , 0
Permanent Ineff=
       F       F
Bank Sta=4985,5015
XS Rating Curve= 0 ,0
Exp/Cntr=0.3,0.1

Type RM Length L Ch R = 1 ,53658   ,85,85,85
BEGIN DESCRIPTION:
Georges Creek 107.7
END DESCRIPTION:
XS GIS Cut Line= 4
      1518716.49       1098356.7      1519014.06      1098084.56
      1519077.65        1097993.      1519118.34      1097809.88
#Sta/Elev= 27
  4533.4  986.01  4565.9   985.2  4610.7  981.87  4625.7  981.38  4643.6  978.86
  4749.9  976.63  4776.4  975.86  4802.2  975.56  4847.7  973.22  4865.9  972.77
  4925.9  971.12  4936.7  970.97  4939.3  970.89  4977.1  966.08  4983.6  962.63
    4989   959.5  4994.5   952.4  5005.5   952.4    5011   959.5  5048.1  966.98
    5117   972.4  5146.1  980.53  5187.2  991.11  5192.5  992.06  5196.7   992.9
  5201.9  992.59  5219.5  992.28
#Mann= 3 ,-1,0
  4533.4    .135       0    4989     .05       0    5011     .15       0
#XS Ineff= 2 , 0
Permanent Ineff=
       F       F
Bank Sta=4989,5011
XS Rating Curve= 0 ,0
Exp/Cntr=0.3,0.1
