HEC-RAS study 12mile_Combined.prj: 12mile Creek Combined Model

--- 12mile_Combined.g01 (geometry) --- (continued)

Type RM Length L Ch R = 1 ,65446.48,304.5831,406.3046,353.6302
XS GIS Cut Line= 3
   1495002.60171   1140238.58005   1494720.80873   1140467.92552
   1494376.79035   1140757.71916
#Sta/Elev= 30
 -364.93 1021.33 -353.67 1017.08 -322.36 1012.31 -307.28 1008.27 -296.23 1006.95
 -284.79 1007.13 -238.77  996.83 -157.87  990.22 -108.02  989.85  -94.08   990.8
  -42.05  988.63  -14.31  990.11   -5.62  987.09   -2.86  985.66    4.88  987.15
    6.89  989.28    8.27  989.41   26.38988.6756   70.12   990.4  193.44  991.58
  206.65  988.78  214.36  989.49  224.46  993.69  247.88993.1054  281.65  993.97
  295.35  996.11  341.46  997.06  373.99  999.25  395.62  999.05  448.21 1002.72
#Mann= 5 ,-1,0
 -364.93    .135       0   -5.62     .04       0    4.88     .13       0
   26.38      .1       0  247.88     .06       0
Bank Sta=-5.62,4.88
XS Rating Curve= 0 ,0
Exp/Cntr=0.3,0.1

Type RM Length L Ch R = 1 ,65040.18,35.51299,81.20195,61.46384
BEGIN DESCRIPTION:
TWE_34USX
END DESCRIPTION:
XS GIS Cut Line= 4
   1494908.63911   1140071.05282   1494541.28051    1140195.3481
   1494498.83563   1140223.13156   1494204.29757   1140400.56759
#Sta/Elev= 30
 -438.52 1003.72 -401.03  995.42 -363.64  992.64 -342.29  992.77 -244.04  990.21
    -218  990.59 -155.56  989.34 -135.13  990.65 -127.08  989.72  -92.17  988.85
  -44.01  989.12   -8.64  987.83   -5.62  985.59   -2.86  984.16    4.88  985.65
    9.92  987.67   39.94  987.44   99.12  988.58  182.89  988.58  185.38  988.03
  196.63  986.58  202.87  989.31  205.73  989.72  235.33  991.68  269.95  996.14
  295.21 1000.97  304.43 1001.98  313.04 1005.83  326.54  1006.6  343.89 1011.02
#Mann= 6 ,-1,0
 -438.52    .135       0   -5.62     .04       0    4.88     .13       0
   39.94      .1       0  185.38     .14       0  326.54      .1       0
#XS Ineff= 2 , 0
         -265.47  993.63   178.9          993.91
Permanent Ineff=
       F       F
Bank Sta=-5.62,4.88
XS Rating Curve= 0 ,0
Exp/Cntr=0.5,0.3

Type RM Length L Ch R = 1 ,64958.98,48.1625,49.4349,49.77205
BEGIN DESCRIPTION:
Tater Hill Mountain Rd (TWE_34) - US
END DESCRIPTION:
XS GIS Cut Line= 3
   1494928.16207   1140005.96654     1494427.646   1140206.32808
   1494156.11417   1140313.08399
#Sta/Elev= 30
 -541.18 1005.67 -514.07   999.8 -479.72  994.75 -450.79  992.95 -397.13  991.24
 -365.78  991.73 -300.71  989.91 -117.99  988.77  -97.96  989.43   -52.3  987.22
  -25.54  988.33   -7.99  986.24    -.26  984.62    2.21  983.05    5.39  983.32
    7.94  985.93   10.58  987.28   41.61  988.55   50.38  990.56    56.2  990.84
  122.18   991.2  176.14  993.16  189.09  994.68  225.34 1001.58  239.97 1001.94
  247.04 1004.24  255.82 1004.98  266.81 1003.89  276.66 1003.95  289.72 1006.92
#Mann= 6 ,-1,0
 -541.18    .135       0   -52.3      .1       0   -7.99     .04       0
    7.94      .1       0  122.18     .14       0  266.81      .1       0
#XS Ineff= 2 , 0
       0     -30     989      20       0     992
Permanent Ineff=
       F       F
Bank Sta=-7.99,7.94
XS Rating Curve= 0 ,0
Exp/Cntr=0.5,0.3

Type RM Length L Ch R = 3 ,64934.13,,,
BEGIN DESCRIPTION:
Tater Hill Mountain Rd (TWE_34) - TOR
END DESCRIPTION:
Bridge Culvert--1,0,-1,-1, 0
Deck Dist Width WeirC Skew NumUp NumDn MinLoCord MaxHiCord MaxSubmerge Is_Ogee
11.15,27.4,2.6,0, 96, 96, 989.34, , 0.95, 0, 0,0,,
 -546.76 -545.95  -545.1 -544.55 -544.05 -542.39  -540.6 -539.85 -538.13 -537.16
 -535.26 -532.87 -529.52 -529.28 -527.52 -525.34 -523.28    -489 -473.84 -454.19
 -430.41 -427.48 -419.64 -413.23 -406.36 -397.13 -389.85 -385.12 -375.47 -356.87
 -347.12 -343.48  -334.6 -327.55 -320.63 -310.81 -297.34 -285.71 -243.43  -217.8
 -191.58    -165 -139.38 -114.76  -87.68  -61.89  -19.41  -19.41  -17.41  -17.41
    8.57    8.57   10.27   10.27   10.55   47.67   71.34   89.86   120.5  146.19
  172.99  199.51  207.88  226.01  250.95  251.15  253.29  253.59  254.64  255.29
  256.14  257.54  259.25  261.16  262.55  264.78  265.26  266.61  269.54  271.23
   273.1  273.44  273.94  276.27  276.34   276.4  278.63  279.39  280.85  283.71
  284.18  286.24  287.66  288.87  289.67  289.92
 1004.41 1004.29 1004.11 1004.07 1003.99  1003.7 1003.32 1003.21 1003.05 1002.86
 1002.58 1002.24 1001.61 1001.56 1001.32 1000.99 1000.57  995.29  993.67  993.12
   992.7  992.66  992.54   992.4  992.24  992.06   991.9  991.81   991.6   991.3
  991.24  991.15  991.05  990.97  990.95  990.87   990.7  990.63  990.26  990.18
     990  989.51  989.34  989.52  989.45  989.87  990.77   993.5   993.5   993.5
   994.2   994.2   994.2   991.5   991.5  992.07  992.76  993.54  994.83   996.3
   997.8  999.92 1000.58 1002.01 1003.96 1003.56 1003.79 1003.81 1003.81 1003.82
 1003.91 1003.99 1004.18 1004.35 1004.46  1004.7 1004.74  1004.8 1005.03 1005.22
 1005.39 1005.42 1005.52 1005.74 1005.74 1005.75 1005.96 1005.97 1006.08 1006.34
 1006.39 1006.61  1006.8 1006.93 1006.94 1006.95
                                                                                
                                                                                
                                                                                
                                                                                
                                                                          989.36
     990
                                                                                
                                                                                
                                                                                
                                                
 -546.76 -545.95  -545.1 -544.55 -544.05 -542.39  -540.6 -539.85 -538.13 -537.16
 -535.26 -532.87 -529.52 -529.28 -527.52 -525.34 -523.28    -489 -473.84 -454.19
 -430.41 -427.48 -419.64 -413.23 -406.36 -397.13 -389.85 -385.12 -375.47 -356.87
 -347.12 -343.48  -334.6 -327.55 -320.63 -310.81 -297.34 -285.71 -243.43  -217.8
 -191.58    -165 -139.38 -114.76  -87.68  -61.89  -19.41  -19.41  -17.41  -17.41
    8.57    8.57   10.27   10.27   10.55   47.67   71.34   89.86   120.5  146.19
  172.99  199.51  207.88  226.01  250.95  251.15  253.29  253.59  254.64  255.29
  256.14  257.54  259.25  261.16  262.55  264.78  265.26  266.61  269.54  271.23
   273.1  273.44  273.94  276.27  276.34   276.4  278.63  279.39  280.85  283.71
  284.18  286.24  287.66  288.87  289.67  289.92
 1004.41 1004.29 1004.11 1004.07 1003.99  1003.7 1003.32 1003.21 1003.05 1002.86
 1002.58 1002.24 1001.61 1001.56 1001.32 1000.99 1000.57  995.29  993.67  993.12
   992.7  992.66  992.54   992.4  992.24  992.06   991.9  991.81   991.6   991.3
  991.24  991.15  991.05  990.97  990.95  990.87   990.7  990.63  990.26  990.18
     990  989.51  989.34  989.52  989.45  989.87  990.77   993.5   993.5   993.5
   994.2   994.2   994.2   991.5   991.5  992.07  992.76  993.54  994.83   996.3
   997.8  999.92 1000.58 1002.01 1003.96 1003.56 1003.79 1003.81 1003.81 1003.82
 1003.91 1003.99 1004.18 1004.35 1004.46  1004.7 1004.74  1004.8 1005.03 1005.22
 1005.39 1005.42 1005.52 1005.74 1005.74 1005.75 1005.96 1005.97 1006.08 1006.34
 1006.39 1006.61  1006.8 1006.93 1006.94 1006.95
                                                                                
                                                                                
                                                                                
                                                                                
                                                                          989.36
     990
                                                                                
                                                                                
                                                                                
                                                
BR Coef=-1 , 1 , 0 ,, 0 ,,,0.8,0,1.2,0,
WSPro=,,,, 1 ,,,, 0 ,,,, 0 ,,,,-1 ,-1 ,-1 , 0 , 0 , 0 , 0 , 0
BC Design=,, 0 ,, 0 ,,,,,,
BC Use User HTab Curves=0
BC User HTab FreeFlow(D)= 0

Type RM Length L Ch R = 1 ,64909.54,244.0514,350.0783,339.4108
BEGIN DESCRIPTION:
Tater Hill Mountain Rd (TWE_34) - DS
END DESCRIPTION:
XS GIS Cut Line= 3
    1494916.5584   1139960.32448    1494408.3061   1140161.45932
   1494136.00066   1140265.89469
#Sta/Elev= 30
 -548.25 1003.22 -500.14  995.78 -490.78  993.36 -474.72  993.46 -448.03  992.32
 -423.28  991.73 -356.03  989.53  -74.77  987.93  -28.72  989.12   -19.5   988.1
   -7.99  988.28    -.26  986.66    2.21  985.09    5.39  985.36    7.83  987.94
    8.73     988   20.54  989.56   67.22  991.67   89.74  991.85  109.53  993.41
  150.11  994.86  179.98  997.53  197.28 1000.15  206.36 1003.17  227.54 1006.09
  249.09  1008.4  254.35 1007.86  279.38 1010.73   286.4 1009.95     290 1011.01
#Mann= 7 ,-1,0
 -548.25    .135       0 -474.72     .06       0 -448.03     .06       0
 -423.28      .1       0  -74.77     .13       0   -7.99     .04       0
    8.73     .13       0
#XS Ineff= 2 , 0
       0     -30     989      20       0     992
Permanent Ineff=
       F       F
Bank Sta=-7.99,8.73
XS Rating Curve= 0 ,0
Exp/Cntr=0.5,0.3

Type RM Length L Ch R = 1 ,64559.46,326.2435,338.1874,332.4392
XS GIS Cut Line= 3
   1494955.51411   1139886.15682   1494446.39829   1139848.39633
   1494140.40814   1139821.05217
#Sta/Elev= 30
  -512.4 1014.05 -504.11 1011.43 -492.78 1009.88  -455.3 1001.43 -434.64  994.46
 -425.37995.0964  -413.2  994.78 -403.95993.4351 -376.61  990.15 -331.21  988.57
 -138.39  986.51  -99.19  987.61  -86.37  986.86   -47.1987.0467  -21.81  987.68
    -8.9  986.85   -7.92  986.02   -5.86  983.81   -3.59   983.8    6.57  984.13
    9.25  985.78   25.56   987.4  105.07  986.64   183.5  986.69  192.67  987.45
  200.68  993.63   204.1  995.26  244.33 1009.38  276.11 1016.99  305.33 1021.81
#Mann= 6 ,-1,0
  -512.4    .135       0 -425.37     .06       0 -403.95      .1       0
   -47.1    .135       0   -7.92     .04       0    9.25    .135       0
Bank Sta=-7.92,9.25
XS Rating Curve= 0 ,0
Exp/Cntr=0.3,0.1

Type RM Length L Ch R = 1 ,64221.28,399.8014,479.3083,372.4897
XS GIS Cut Line= 3
   1494915.14928   1139558.03117   1494480.25262   1139524.17684
    1494308.3773    1139518.9685
#Sta/Elev= 30
 -439.77 1021.03 -399.69 1006.19  -387.7998.5498 -386.14  997.55 -376.76  998.54
    -368  998.44 -361.45996.7295  -357.7  995.15 -353.88  995.08  -342.3  992.06
 -322.42990.6046 -233.05  987.25 -150.52986.0724  -60.55  985.42    -9.9  985.87
   -7.92  984.22   -5.86982.0099   -3.59     982    6.57  982.33    9.25  983.98
   14.41  985.69   29.87  986.15   37.35  989.91    45.5  995.43   49.85  999.45
   53.19 1000.87   61.45 1006.65   79.86 1011.73  102.39 1014.93   168.4 1019.33
#Mann= 7 ,-1,0
 -439.77    .135       0  -387.7     .06       0 -361.45     .14       0
 -322.42      .1       0 -150.52    .135       0   -7.92     .04       0
    9.25    .135       0
Bank Sta=-7.92,9.25
XS Rating Curve= 0 ,0
Exp/Cntr=0.3,0.1

Type RM Length L Ch R = 1 ,63741.97,414.8988,535.5957,451.0252
XS GIS Cut Line= 3
   1494924.26411   1139068.44685   1494457.15322   1139147.25558
   1494060.98097   1139215.58268
#Sta/Elev= 30
 -475.64 1006.63 -425.01   998.8 -409.71  994.22 -389.08  993.57  -379.4  990.61
 -349.35987.1844 -309.01  986.27 -279.99  984.66 -209.88984.4842 -151.29  984.54
 -145.71  985.44 -115.67  985.15 -103.69  984.35  -75.35  985.52  -58.78  984.23
  -39.85  985.06   -17.6  984.58    -8.9   983.1   -7.92  982.27   -5.86  980.06
   -3.59  980.05    6.57  980.38    9.25  982.03   11.61  984.73   88.69984.5318
   157.4  984.68  180.78  986.01  266.03  987.21  366.89  992.05   400.1  995.02
#Mann= 6 ,-1,0
 -475.64     .11       0 -349.35     .14       0 -209.88     .12       0
   -7.92     .04       0    9.25     .12       0   88.69     .13       0
#XS Ineff= 1 ,-1
  179.65  295.77  988.05
Permanent Ineff=
       F
Bank Sta=-7.92,9.25
XS Rating Curve= 0 ,0
Exp/Cntr=0.3,0.1

Type RM Length L Ch R = 1 ,63206.37,683.8718,710.6496,611.7475
BEGIN DESCRIPTION:
TWE_33X
END DESCRIPTION:
XS GIS Cut Line= 5
   1494752.55512    1138692.6063   1494461.53675   1138724.07907
   1494396.40617   1138716.21424   1494327.71129   1138708.10335
    1494165.5315   1138691.52133
#Sta/Elev= 30
 -358.32 1026.38 -342.77 1021.55 -290.65 1001.71 -282.43  994.42 -279.93  993.14
 -276.56  992.44 -262.46  992.81 -257.93  991.64 -254.67  989.53 -241.47  985.36
 -229.09  983.18 -169.67  982.67    -130  983.53 -124.37  982.64  -25.97  982.66
  -13.47  982.13   -7.92  979.81   -5.86   977.6   -3.59  977.59    6.57  977.92
    9.25  979.57   14.72  981.99    28.2   982.8  123.71  987.46  128.01  988.01
  149.03  995.42  157.77  996.68  191.79  998.37  223.47 1002.05  232.19 1002.22
#Mann= 5 ,-1,0
 -358.32     .14       0 -254.67     .12       0   -7.92     .04       0
    9.25     .12       0    28.2     .12       0
Bank Sta=-7.92,9.25
XS Rating Curve= 0 ,0
Exp/Cntr=0.3,0.1

Type RM Length L Ch R = 1 ,62495.72,535.3537,586.2144,526.637
XS GIS Cut Line= 3
   1494925.29856   1137786.57152   1494243.00558   1138119.90551
   1493998.21325   1138224.07251
#Sta/Elev= 30
 -764.85 1009.08 -714.35 1001.51  -653.5  995.12 -636.71  992.47 -598.27  988.32
 -581.37  987.71  -559.1   985.7 -546.46  985.47 -532.98  983.84 -517.08  984.21
  -447.1  982.76 -365.55  982.32 -288.16  980.77 -170.05980.1938 -129.68   979.8
  -21.24  980.43   -9.61  979.76   -6.34  975.54     .01   975.1    7.93  977.63
    9.21  979.51    23.5  980.32   31.22   981.5   79.59  983.76   85.72  983.43
  179.89  990.26  188.63   991.7   206.3  996.09  253.64 1000.86  260.55 1002.47
#Mann= 4 ,-1,0
 -764.85     .14       0 -170.05     .12       0   -9.61     .04       0
    9.21     .14       0
#XS Ineff= 2 ,-1
 -543.98 -516.77  984.21 -494.19 -437.29  983.36
Permanent Ineff=
       F       F
Bank Sta=-9.61,9.21
XS Rating Curve= 0 ,0
Exp/Cntr=0.3,0.1

Type RM Length L Ch R = 1 ,61909.51,384.125,546.4482,467.8672
XS GIS Cut Line= 3
   1494607.58957   1137362.09154   1494103.69948   1137612.11844
   1493912.27592   1137708.44619
#Sta/Elev= 30
 -559.24 1013.74 -526.83 1003.95 -497.91  997.17 -477.85  995.62 -463.52  991.18
 -438.23  986.66 -428.06  983.99 -399.87  980.11 -277.65   978.8  -258.3  979.38
 -125.01978.5942  -44.54  979.49  -23.91  978.57  -17.78  979.28   -9.61  977.76
   -6.34  973.54     .01   973.1    7.93  975.63    9.21  977.51   10.07  979.17
   12.25   979.3   39.03978.7529    76.2  979.19   93.02  987.88  105.51   990.5
  115.93  999.49  120.42 1001.46   132.7 1003.19   154.21004.242  217.56 1008.05
#Mann= 6 ,-1,0
 -559.24     .14       0 -125.01     .12       0   -9.61     .04       0
    9.21     .12       0   39.03     .14       0   154.2      .1       0
Bank Sta=-9.61,9.21
XS Rating Curve= 0 ,0
Exp/Cntr=0.3,0.1

Type RM Length L Ch R = 1 ,61363.06,113.0541,47.42634,15.37912
BEGIN DESCRIPTION:
TWE_32USX
END DESCRIPTION:
XS GIS Cut Line= 6
   1494472.47474   1137136.85072   1494079.67881   1137171.57316
   1493944.05184   1137176.11975   1493876.87697   1137238.33924
   1493843.28904   1137330.29199   1493842.18799   1137503.73556
#Sta/Elev= 30
 -479.03  995.53 -457.36  991.76 -403.83   987.1  -306.1  982.57 -123.74   977.5
  -44.04  976.51     -40  973.81  -32.47  972.68  -27.62  973.43   -26.1  976.36
   -9.61  976.03   -6.34  971.81     .01  971.37    7.93   973.9    9.21  975.78
    20.2  976.99  101.28  977.89  129.32  982.65  142.79  987.45  161.77  989.28
  174.39  987.62  187.34  988.09  192.88  986.42  230.07  990.16  251.72  988.37
  270.79  996.75  287.91   997.8  296.84  997.01  338.71  997.88  413.94 1002.94
#Mann= 6 ,-1,0
 -479.03     .14       0 -123.74     .12       0  -44.04    .045       0
   -26.1     .12       0   -9.61     .04       0    9.21     .12       0
Bank Sta=-9.61,9.21
XS Rating Curve= 0 ,0
Exp/Cntr=0.5,0.3

Type RM Length L Ch R = 1 ,61315.64,58.08566,71.82238,65.56407
BEGIN DESCRIPTION:
Ponderosa Rd (TWE_32) - US
END DESCRIPTION:
XS GIS Cut Line= 6
   1494370.79232   1136888.40617   1493919.27428   1137183.82841
   1493869.16831   1137236.13681   1493848.24475   1137276.33169
   1493831.72638   1137341.30413    1493831.7792   1137482.21719
#Sta/Elev= 30
 -361.86 1000.19-339.301  990.74-334.706  989.52-323.516  988.71 -274.08  987.31
-263.472  984.82-242.854  982.45-238.021   981.9 -228.06  982.78-219.082  981.55
-200.193  983.23-192.927  980.79-176.855  982.04-172.735  980.87-164.527  980.37
-157.023  978.34  -63.46  977.05 -10.887  976.72  -7.176  971.63  -2.818  971.13
   7.888  973.53  10.526  976.48   97.79  977.72 126.526  983.15  136.34  986.43
 212.185   991.9 234.015   992.7 264.807  996.52 305.208  999.35 346.935 1002.44
#Mann= 7 ,-1,0
 -361.86     .14       0-323.516     .11       0-242.854     .14       0
  -63.46     .12       0 -10.887     .04       0  10.526     .12       0
 305.208     .06       0
#XS Ineff= 3 ,-1
 -361.86 -200.19     985     -39    -200   980.5      35 346.935   980.5
Permanent Ineff=
       F       F       F
Bank Sta=-10.887,10.526
XS Rating Curve= 0 ,0
Skew Angle= 35
Exp/Cntr=0.5,0.3

Type RM Length L Ch R = 3 ,61281.73,,,
BEGIN DESCRIPTION:
Ponderosa Rd (TWE_32) - TOR
Skew = 35 Degrees
END DESCRIPTION:
Bridge Culvert--1,0,-1,-1, 0
Deck Dist Width WeirC Skew NumUp NumDn MinLoCord MaxHiCord MaxSubmerge Is_Ogee
20,27.5,2.6,35, 169, 169, 980.35, , 0.95, 0, 0,0,,
-362.065-348.852-348.344-344.912-338.875-337.474 -335.14-332.289-329.463-328.341
-326.104-317.307-316.946-313.702-312.015-308.517-304.028-303.234 -301.03-300.932
-300.817-297.909-295.992-293.011-289.832 -286.13-281.469-280.355-279.544-277.906
-276.308-268.641-268.125-267.797-252.217-215.863-213.135-196.441-175.987-154.869
-134.578-129.221-111.446  -90.23 -69.292 -48.649 -23.977 -23.977 -19.471 -19.471
  15.924  15.924   20.02   20.02  52.557  73.404   93.26  96.996 115.074 133.948
 140.992 164.289 190.608 200.143 226.274 254.232 255.715 255.928 256.051 259.425
 260.466 260.777 262.006  265.52 267.805 269.419 272.393  272.95 274.105 274.768
 277.594 278.888 279.699 282.689 285.089 286.113 288.358 288.997 291.594 294.272
  296.05   297.5 298.499 299.203 300.916 301.923 302.521 303.201 304.913 305.667
 306.076 310.721  311.36 312.662 314.161 314.497 315.447 317.643 318.675 320.837
  321.14 323.844 324.859 326.825 327.276 328.783 332.469 332.838 333.067 334.992
 336.082 337.302 339.948 341.029 342.651 342.848 342.897 343.077  344.74 345.764
 346.485 347.304 349.901  350.63 350.982 352.465 352.579 353.071 353.407 354.947
 355.717 356.241 356.405 358.101 359.796 360.271 360.558 361.877 362.655 363.982
 365.448 365.973 366.366 367.062 368.356 369.028 370.265 370.765  372.19 373.836
  374.23 374.271 374.787 377.547 377.785 379.153 379.472  379.53 379.915
 1002.89 1002.75 1002.55  1001.2  998.68  998.01  996.62  995.47  994.14  993.66
  992.76  989.78  989.67  988.82  988.65   987.9  987.03  986.83  986.48  986.47
  986.45   986.2  986.06   985.9  985.98  986.12  985.74  985.78  985.81  985.91
  985.93  985.89  985.88  985.93  985.58  984.43  984.39  984.12  983.38  982.59
  982.07  981.99  981.74  981.51  981.22  981.01  980.64  983.55  983.55  983.55
  983.26  983.26  983.26  980.35  981.12  981.24  981.49  981.63  982.29  984.07
  984.68  986.69  989.09   989.9  992.13  994.46  994.52  994.54  994.55  994.79
  995.16  995.24  995.26  995.32  995.47  995.56  996.14  996.19  996.19  995.99
   996.1  996.12  996.23  996.45  996.62  996.68  996.76  996.78  997.03  997.08
  997.26  997.35  997.42  997.46  997.73  997.84  997.82  997.81  997.84  997.95
  997.93  998.19  998.23  998.32  998.41  998.44  998.48  998.57  998.67  998.86
  998.87  999.01  999.07   999.2  999.22  999.27  999.54  999.57  999.58  999.74
  999.82   999.9 1000.01 1000.12 1000.16 1000.16 1000.16 1000.19 1000.39 1000.44
 1000.47 1000.51 1000.65 1000.71 1000.74 1000.86 1000.87  1000.9 1000.88 1001.03
 1001.09 1001.12 1001.13  1001.2 1001.35 1001.39 1001.41 1001.44 1001.47 1001.56
 1001.63 1001.66 1001.69 1001.75 1001.89 1001.92 1002.02 1002.04 1002.12 1002.28
 1002.32 1002.32 1002.34 1002.39  1002.4 1002.57  1002.6  1002.6 1002.62
                                                                                
                                                                                
                                                                                
                                                                                
                                                                          979.61
  979.63
                                                                                
                                                                                
                                                                                
                                                                                
                                                                                
                                                                                
                                                                                
                                                                                
                                                                                
                                                                                
                                                                        
 -349.18-348.852-348.344-344.912-338.875-337.474 -335.14-332.289-329.463-328.341
-326.104-317.307-316.946-313.702-312.015-308.517-304.028-303.234 -301.03-300.932
-300.817-297.909-295.992-293.011-289.832 -286.13-281.469-280.355-279.544-277.906
-276.308-268.641-268.125-267.797-252.217-215.863-213.135-196.441-175.987-154.869
-134.578-129.221-111.446  -90.23 -69.292 -48.649 -23.977 -23.977 -19.471 -19.471
  15.924  15.924   20.02   20.02  52.557  73.404   93.26  96.996 115.074 133.948
 140.992 164.289 190.608 200.143 226.274 254.232 255.715 255.928 256.051 259.425
 260.466 260.777 262.006  265.52 267.805 269.419 272.393  272.95 274.105 274.768
 277.594 278.888 279.699 282.689 285.089 286.113 288.358 288.997 291.594 294.272
  296.05   297.5 298.499 299.203 300.916 301.923 302.521 303.201 304.913 305.667
 306.076 310.721  311.36 312.662 314.161 314.497 315.447 317.643 318.675 320.837
  321.14 323.844 324.859 326.825 327.276 328.783 332.469 332.838 333.067 334.992
 336.082 337.302 339.948 341.029 342.651 342.848 342.897 343.077  344.74 345.764
 346.485 347.304 349.901  350.63 350.982 352.465 352.579 353.071 353.407 354.947
 355.717 356.241 356.405 358.101 359.796 360.271 360.558 361.877 362.655 363.982
 365.448 365.973 366.366 367.062 368.356 369.028 370.265 370.765  372.19 373.836
  374.23 374.271 374.787 377.547 377.785 379.153 379.472  379.53 379.915
 1002.89 1002.75 1002.55  1001.2  998.68  998.01  996.62  995.47  994.14  993.66
  992.76  989.78  989.67  988.82  988.65   987.9  987.03  986.83  986.48  986.47
  986.45   986.2  986.06   985.9  985.98  986.12  985.74  985.78  985.81  985.91
  985.93  985.89  985.88  985.93  985.58  984.43  984.39  984.12  983.38  982.59
  982.07  981.99  981.74  981.51  981.22  981.01  980.64  983.55  983.55  983.55
  983.26  983.26  983.26  980.35  981.12  981.24  981.49  981.63  982.29  984.07
  984.68  986.69  989.09   989.9  992.13  994.46  994.52  994.54  994.55  994.79
  995.16  995.24  995.26  995.32  995.47  995.56  996.14  996.19  996.19  995.99
   996.1  996.12  996.23  996.45  996.62  996.68  996.76  996.78  997.03  997.08
  997.26  997.35  997.42  997.46  997.73  997.84  997.82  997.81  997.84  997.95
  997.93  998.19  998.23  998.32  998.41  998.44  998.48  998.57  998.67  998.86
  998.87  999.01  999.07   999.2  999.22  999.27  999.54  999.57  999.58  999.74
  999.82   999.9 1000.01 1000.12 1000.16 1000.16 1000.16 1000.19 1000.39 1000.44
 1000.47 1000.51 1000.65 1000.71 1000.74 1000.86 1000.87  1000.9 1000.88 1001.03
 1001.09 1001.12 1001.13  1001.2 1001.35 1001.39 1001.41 1001.44 1001.47 1001.56
 1001.63 1001.66 1001.69 1001.75 1001.89 1001.92 1002.02 1002.04 1002.12 1002.28
 1002.32 1002.32 1002.34 1002.39  1002.4 1002.57  1002.6  1002.6 1002.62
                                                                                
                                                                                
                                                                                
                                                                                
                                                                          979.63
   979.6
                                                                                
                                                                                
                                                                                
                                                                                
                                                                                
                                                                                
                                                                                
                                                                                
                                                                                
                                                                                
                                                                        
Pier Skew, UpSta & Num, DnSta & Num=  ,-8.814, 4 ,-8.814, 4 , 3 , 3 , 0 ,,
       1       1     1.5     1.5
     970  978.61  978.61     980
       1       1     1.5     1.5
     970  978.61  978.61     980
Pier Skew, UpSta & Num, DnSta & Num=  ,4.751, 4 ,4.751, 4 , 3 , 3 , 0 ,,
       1       1     1.5     1.5
     970  978.61  978.61     980
       1       1     1.5     1.5
     970  978.61  978.61     980
BR Coef=-1 , 1 , 0 ,, 0 ,,,0.8,0,1.2,0,
WSPro=,,,, 1 ,,,, 0 ,,,, 0 ,,,,-1 ,-1 ,-1 , 0 , 0 , 0 , 0 , 0
BC Design=,, 0 ,, 0 ,,,,,,
BC Use User HTab Curves=0
BC User HTab FreeFlow(D)= 0

Type RM Length L Ch R = 1 ,61243.81,387.1822,406.8167,383.6989
BEGIN DESCRIPTION:
Ponderosa Rd (TWE_32) - DS
END DESCRIPTION:
XS GIS Cut Line= 6
   1494339.90584    1136838.5899   1493913.69751   1137112.57776
   1493841.74245    1137191.2897   1493809.85991   1137248.08038
   1493783.95538   1137353.69094   1493788.93701   1137476.23917
#Sta/Elev= 30
 -331.92 1005.25-313.023  996.41 -293.15     989-281.018  986.59-241.363  986.09
-211.472  983.93-189.929  981.98-130.114  980.31-106.908  977.67   -87.1  977.18
 -11.747  976.62 -10.887  973.43  -7.176  968.34  -2.818  967.84   7.888  970.24
  10.526  973.19  18.152  976.53 118.204  976.87 142.901  979.11 149.299  980.72
 172.341  986.65 190.756  988.41 219.844  994.37 237.906  993.02 253.052  993.48
 259.851  994.01 274.719  997.72 357.429 1001.41 389.441 1004.42 413.565 1004.93
#Mann= 9 ,-1,0
 -331.92     .14       0 -293.15     .11       0-241.363     .06       0
-211.472     .14       0   -87.1     .12       0 -10.887     .04       0
  10.526     .12       0 149.299      .1       0 389.441     .14       0
#XS Ineff= 2 , 0
       0     -40   980.5      35       0   980.5
Permanent Ineff=
       F       F
Bank Sta=-10.887,10.526
XS Rating Curve= 0 ,0
Skew Angle= 35
Exp/Cntr=0.5,0.3

Type RM Length L Ch R = 1 ,60836.99,650.8298,841.0577,674.1644
XS GIS Cut Line= 3
   1494205.80315   1136466.79462   1493779.22999   1136747.10105
   1493416.13419   1136988.72146
#Sta/Elev= 30
 -509.67    1013  -499.5 1010.85 -470.69 1002.15  -457.8  994.27 -454.15  993.24
 -446.55  994.02 -431.96  993.44 -419.85  989.82 -409.21  987.88 -389.36   986.3
 -376.77  982.59 -366.88  981.19 -247.38  976.35 -196.38  975.79 -104.25  974.89
  -22.06  975.57   -17.3  975.06  -16.12  974.02  -14.93  972.34    5.12   971.5
   18.08  972.83   21.34  975.34   79.56  973.93  193.47  974.74  236.31  974.95
   311.1  982.06     338  983.89  365.44  987.55  386.81  988.63   436.9  993.95
#Mann= 9 ,-1,0
 -509.67     .14       0 -446.55     .06       0 -419.85     .14       0
 -196.38     .12       0  -16.12     .04       0   18.08     .12       0
  193.47     .12       0  236.31     .14       0   311.1      .1       0
#XS Ineff= 2 , 0
                          269.36          989.92
Permanent Ineff=
       F       F
Bank Sta=-16.12,18.08
XS Rating Curve= 0 ,0
Exp/Cntr=0.3,0.1

Type RM Length L Ch R = 1 ,59995.94,1016.771,1103.151,955.7007
XS GIS Cut Line= 4
   1493900.16142   1135930.25492   1493450.41831   1136177.14272
   1493236.87631   1136302.14304    1493177.9393   1136958.03281
#Sta/Elev= 30
 -515.04 1010.82 -506.69 1009.11 -499.77  1004.7  -495.1 1005.24  -469.8 1006.13
 -455.61 1007.28 -374.03 1002.98 -345.81 1002.79 -307.22 1000.38 -250.48  994.47
 -169.46  989.53 -143.18   985.9 -104.14  973.96  -98.96  973.71  -77.03  972.16
  -16.12  971.77  -14.93  970.09    5.12  969.25   18.08  970.58   18.53  971.97
  159.77  972.36  170.16   972.9  176.45  975.36  219.16  983.49  281.51  987.56
  338.91  987.03  455.34  980.32  797.21  993.49  833.03  998.17  903.98  999.43
#Mann= 7 ,-1,0
 -515.04     .14       0  -495.1     .06       0  -469.8     .14       0
  -98.96     .12       0  -16.12     .04       0   18.53     .12       0
  159.77     .14       0
#XS Ineff= 2 , 0
                          303.33           996.1
Permanent Ineff=
       F       F
Bank Sta=-16.12,18.53
XS Rating Curve= 0 ,0
Exp/Cntr=0.3,0.1

Type RM Length L Ch R = 1 ,58892.79,585.639,764.8176,605.2095
XS GIS Cut Line= 3
   1493190.86877   1134992.24475   1492643.99278   1135673.66962
   1491849.72047   1136737.04003
#Sta/Elev= 30
 -884.33 1021.41 -795.52 1002.97  -770.5   996.3 -727.55  987.31 -696.76   982.2
 -635.48  976.38 -485.27  971.52 -286.17  968.56  -100.4  968.53  -26.73  969.73
   -16.8  969.48  -16.12  968.52  -14.93  966.84    5.12     966   17.82  967.28
   18.78  968.42   20.36   969.5  168.59  968.18  555.69   969.6   695.7  971.27
  790.66  970.53  882.52   972.1 1021.45  978.05  1085.6  986.61  1118.7  990.65
 1140.68  991.61 1166.86  995.03 1203.34  997.45 1261.21  999.95 1316.67 1000.27
#Mann= 5 ,-1,0
 -884.33     .13       0  -16.12     .04       0   18.78     .13       0
  555.69     .14       0  1085.6      .1       0
#XS Ineff= 2 , 0
                          520.13             992
Permanent Ineff=
       F       F
Bank Sta=-16.12,18.78
XS Rating Curve= 0 ,0
Exp/Cntr=0.3,0.1

Type RM Length L Ch R = 1 ,58127.97,653.5295,1114.794,595.4461
XS GIS Cut Line= 4
   1492709.09744   1134653.70243    1492340.1729   1135122.45341
   1491880.10269   1135678.00984   1491219.16306   1135902.89304
#Sta/Elev= 30
  -615.5 1019.82 -607.64 1019.29 -600.34 1017.31  -593.2 1012.04 -584.65 1008.02
 -563.25 1000.73 -520.19  989.79 -441.42  977.47 -383.41  971.83 -309.46  969.18
 -301.33  966.85 -265.32   965.9  -53.13  966.73  -18.99  966.48  -16.12  965.52
  -14.93  963.84    5.12     963   17.82  964.28   19.09  965.58   20.34  966.53
  271.28  967.41  708.23  966.52  863.57  966.12  924.56  967.28 1228.79   968.4
 1254.58  970.69 1284.75  979.61 1309.18   984.3  1372.7  987.58 1400.49  987.21
#Mann= 4 ,-1,0
  -615.5     .13       0  -16.12     .04       0   19.09     .13       0
  708.23     .14       0
#XS Ineff= 2 , 0
                          721.94          996.12
Permanent Ineff=
       F       F
Bank Sta=-16.12,19.09
XS Rating Curve= 0 ,0
Exp/Cntr=0.3,0.1

Type RM Length L Ch R = 1 ,54857.69,50.84569,55.41602,71.15096
BEGIN DESCRIPTION:
Dam E. of Midway RD (TWE_30) - DS
END DESCRIPTION:
XS GIS Cut Line= 6
   1490592.03937   1133108.30348   1490503.49738   1133333.99869
   1490269.14436   1133620.46982   1490107.66339        1133959.
   1490126.76083   1134085.73589   1490404.53904   1134547.54265
#Sta/Elev= 30
 -611.27 1008.93  -606.9 1009.08 -588.71 1002.67 -544.08   992.8 -497.29  987.74
 -457.94  979.16 -442.33  977.69 -263.42   977.8 -247.92  981.25 -169.91  974.56
  -95.72  961.06   -48.4  958.62  -40.16  951.66  -35.39  948.58   -3.66  945.04
   34.33     948   40.07   951.3   51.54  958.15    91.9  959.54  175.84  961.67
  223.66  965.06  359.54  960.82  558.15  962.97  646.16  965.58  704.55  972.37
  742.04  970.43  861.17  978.39  876.49  982.23  900.66   984.9  1050.6  990.99
#Mann= 6 ,-1,0
 -611.27     .14       0 -442.33      .1       0 -263.42     .14       0
  -40.16    .045       0   40.07     .14       0    91.9     .14       0
Bank Sta=-40.16,40.07
XS Rating Curve= 0 ,0
Exp/Cntr=0.5,0.3

Type RM Length L Ch R = 1 ,54802.28,527.0717,693.4466,535.7596
BEGIN DESCRIPTION:
TWE_30DSX
END DESCRIPTION:
XS GIS Cut Line= 6
   1490564.26148   1133103.09514   1490480.92815   1133335.73458
   1490310.07087   1133498.24409   1490226.75427   1133585.52756
   1489909.04528   1133906.70899   1489820.50361   1134158.44554
#Sta/Elev= 30
 -607.24  1005.6 -587.76  996.82 -526.14  985.43 -469.43  979.52 -450.12  981.52
  -438.5     978 -274.69  975.87 -216.89  974.22  -68.13  959.16   -64.6  952.09
  -62.97  948.83  -35.39  949.83   -3.66  946.18   14.12  948.66   48.08  948.55
   52.26  949.45   53.83  952.18   56.22  956.43   65.11  957.73  167.68  958.06
  182.76  954.48   192.7  957.44  204.68  952.58  226.02  957.75  294.47  960.05
  326.94  968.08  378.82  974.22  599.72  975.46  638.16  981.58  714.96  984.85
#Mann= 5 ,-1,0
 -607.24     .14       0  -438.5      .1       0 -274.69     .14       0
   -64.6     .04       0   53.83     .14       0
#XS Ineff= 2 , 0
                          100.27          963.98
Permanent Ineff=
       F       F
Bank Sta=-64.6,53.83
XS Rating Curve= 0 ,0
Exp/Cntr=0.3,0.1

Type RM Length L Ch R = 1 ,54108.83,630.9732,650.1635,610.911
XS GIS Cut Line= 4
   1490429.87992   1132957.27165   1490076.14665   1133111.35138
   1489466.75131   1133383.54823   1489171.19685   1133373.93898
#Sta/Elev= 30
 -392.97  985.58 -361.18  975.01  -342.1  971.15  -326.9  971.15 -299.64  967.61
 -286.73  964.16 -241.56  958.92   -85.3  954.16  -42.91  955.91  -16.28  954.64
   -13.2  951.46  -11.14  946.33   -7.94  946.12    7.19  947.22   11.26  951.52
   15.95  954.16   60.71955.2551  162.96  954.56   174.7  957.15   186.4  957.15
  252.22  963.53  279.18   964.5   427.2  960.88  435.43961.8668  461.49960.7619
   466.2  959.34  502.29  959.08  525.06960.9039  868.76  965.89     956  971.79
#Mann= 7 ,-1,0
 -392.97     .14       0   -13.2     .04       0   11.26     .14       0
   60.71     .12       0  435.43     .06       0  461.49      .1       0
  525.06     .14       0
Bank Sta=-13.2,11.26
XS Rating Curve= 0 ,0
Exp/Cntr=0.3,0.1

Type RM Length L Ch R = 1 ,53458.67,464.3838,527.3426,535.4126
BEGIN DESCRIPTION:
TWE_29X
END DESCRIPTION:
XS GIS Cut Line= 5
    1490097.8481    1132375.6729   1489884.26542   1132511.71916
   1489794.05807   1132565.68701   1489741.91503    1132599.0584
   1489425.10367   1132670.81266
#Sta/Elev= 30
 -358.57  982.99 -325.85  978.92 -282.67  970.98 -244.38  955.07 -221.78  953.27
 -192.62  953.26 -120.13  953.38  -75.94  952.52  -24.52  953.83  -16.28  953.74
   -13.2  950.56  -11.14  945.43   -7.94  945.22    7.19  946.32   11.26  950.62
   15.95  953.26   47.39  952.87   94.28  953.03   112.7  953.11  132.78  954.35
  171.45  958.68  189.16  959.21  204.42  961.22  212.93  961.45   232.2  959.98
  236.63   961.2  240.46  963.16  253.86  966.24  283.97  967.79  386.52  972.86
#Mann= 10 ,-1,0
 -358.57    .135       0 -192.62      .1       0  -24.52     .12       0
   -13.2     .04       0   11.26      .1       0   47.39     .12       0
   94.28      .1       0  212.93     .06       0  236.63      .1       0
  283.97     .14       0
#Block Obstruct= 1 ,-1
     130     160     960
Bank Sta=-13.2,11.26
XS Rating Curve= 0 ,0
Exp/Cntr=0.3,0.1

Type RM Length L Ch R = 1 ,52931.33,302.7447,311.809,300.2909
XS GIS Cut Line= 3
   1489967.63944   1132024.10991   1489550.97178   1132110.91535
   1489288.38484   1132173.84974
#Sta/Elev= 30
 -428.46  985.79  -389.8  976.98 -361.73   969.6  -312.1   953.8 -286.96952.1042
 -137.06  950.93  -80.65   952.4  -22.76  952.23  -18.38   951.8  -10.93  948.18
   -6.18  943.73    3.41  945.04    6.37  946.18    8.04  947.95    9.87  948.02
   14.92  951.74   18.53  953.11   24.77 953.114   32.25  952.65   73.47  953.51
  124.34  956.34  137.95 960.172  153.09  960.31  167.34   959.2  171.89961.4764
  182.59  965.87  224.74  971.28  243.83  975.28  255.92  977.01  267.17  979.82
#Mann= 7 ,-1,0
 -428.46    .135       0 -286.96      .1       0  -10.93     .04       0
    8.04     .12       0   24.77      .1       0  137.95     .06       0
  171.89     .14       0
Bank Sta=-10.93,8.04
XS Rating Curve= 0 ,0
Exp/Cntr=0.3,0.1

Type RM Length L Ch R = 1 ,52619.52,161.9004,84.63351,63.53086
BEGIN DESCRIPTION:
TWE_28USX
END DESCRIPTION:
XS GIS Cut Line= 5
   1489938.41207   1131819.97211   1489761.47966   1131763.87139
   1489479.48983   1131817.76739   1489378.52165   1131847.61122
   1489280.30938   1131944.04068
#Sta/Elev= 30
 -472.44  990.46 -438.87  987.13 -428.68  985.25 -419.86  982.98 -404.17  977.99
 -388.52  972.34 -356.74  958.66 -352.19  956.88 -347.82  955.78 -339.28  954.14
 -334.91  954.02 -138.03  950.26  -37.33  949.35  -12.53  950.48  -10.93  947.58
   -6.18  943.13    1.74  944.04    6.37  945.58   13.37  947.07   21.09  947.16
   34.36  952.44   44.39  952.09  105.95  953.41  179.19  958.01  192.01  959.16
  213.37  962.37  225.55   964.9  235.42  968.05  238.56  968.23  243.19  968.16
#Mann= 6 ,-1,0
 -472.44    .135       0 -347.82      .1       0  -10.93    .045       0
    6.37     .12       0   44.39      .1       0  238.56     .06       0
Bank Sta=-10.93,6.37
XS Rating Curve= 0 ,0
Exp/Cntr=0.5,0.3

Type RM Length L Ch R = 1 ,52534.89,49.06389,39.87159,41.53906
BEGIN DESCRIPTION:
SE. of Midway RD (TWE_28) - US
END DESCRIPTION:
XS GIS Cut Line= 5
   1489732.33202   1131463.35663   1489607.83694   1131586.93045
   1489447.63845   1131739.82251   1489351.36909   1131838.56037
    1489265.9603   1131927.27625
#Sta/Elev= 30
-399.155  964.63-381.483   962.4-367.805   959.6-347.244  956.91-337.999  956.33
-328.535  954.88-301.209  952.82-268.146  951.78-119.992  950.33 -74.854  949.31
 -44.639  949.81 -21.368  949.17 -16.617  948.14 -11.516  948.18  -7.242  944.61
  -4.573  943.17   -.269  942.63   3.447  944.78   7.661  945.27  12.841  947.98
  17.762  947.65  22.962  949.01  29.786  951.83  40.824  951.47 110.906  953.23
 192.395  957.59 214.969   960.1 245.931  967.94 249.686  968.06 256.251  968.38
#Mann= 6 ,-1,0
-399.155     .13       0-328.535      .1       0 -11.516    .045       0
  12.841     .12       0  40.824      .1       0 249.686     .06       0
#XS Ineff= 2 , 0
       0     -30     950      30       0  951.84
Permanent Ineff=
       F       F
Bank Sta=-11.516,12.841
XS Rating Curve= 0 ,0
Skew Angle= 5
Exp/Cntr=0.5,0.3

Type RM Length L Ch R = 3 ,52513.90,,,
BEGIN DESCRIPTION:
SE. of Midway RD (TWE_28) - TOR
Skew = 5 degrees
END DESCRIPTION:
Bridge Culvert--1,0,-1,-1, 0
Deck Dist Width WeirC Skew NumUp NumDn MinLoCord MaxHiCord MaxSubmerge Is_Ogee
15,12,2.6,5, 88, 88, 950.72, , 0.95, 0, 0,0,,
-394.842-393.078-391.694-391.584-389.482 -387.36-387.281-386.534-385.238-380.566
-380.088-379.889-377.139-372.398 -369.02-368.283-368.214 -366.61-360.702-359.357
-355.203-352.932-349.654-336.764-335.698-335.568-335.379 -332.42-331.803-331.155
-324.779-323.972-323.684-322.309-319.041-310.285-295.471-278.885-260.804-252.167
-244.008-238.369 -227.82-207.378 -178.04-177.293-150.336-120.908 -93.104 -67.393
  -41.93 -15.292 -15.292 -13.797 -13.797  12.851  12.851  14.345  14.345  33.183
  50.208  67.034   89.01 111.863 139.487 171.804 198.831 224.473 227.939 229.444
  230.36 236.068 236.357 236.536 236.676 240.163 245.064 245.821 247.843 249.696
 253.263 254.827 255.942 257.108 259.628 260.057 261.202 261.312
  965.61  965.48   965.2  965.17  964.82  964.33  964.31  964.15  963.82  962.67
  962.55   962.5  961.81  960.86  960.06  959.79  959.77  959.54  958.76  958.49
  957.97  957.72  957.32  955.72   955.6  955.58  955.56  955.24  955.18  955.13
  954.63  954.57  954.55  954.49  954.32  953.81  953.09  952.66  952.26  952.08
  951.99  951.92  951.78   951.7  951.37  951.36  951.11  950.86  950.72  950.97
  951.58  951.75  952.75  952.75  952.75  952.99  952.99  952.99  952.01  952.54
  952.81     953  953.38  954.12  954.95   956.6  958.81  962.92  963.24  963.65
  963.86  964.99  965.04  965.09  965.11   965.8  966.85     967   967.4  967.76
  968.26  968.46  968.49  968.53  968.52  968.56  968.53  968.52
                                                                                
                                                                                
                                                                                
                                                                                
                                                                                
                                  950.13   950.4
                                                                                
                                                                                
                                                                
-394.842-393.078-391.694-391.584-389.482 -387.36-387.281-386.534-385.238-380.566
-380.088-379.889-377.139-372.398 -369.02-368.283-368.214 -366.61-360.702-359.357
-355.203-352.932-349.654-336.764-335.698-335.568-335.379 -332.42-331.803-331.155
-324.779-323.972-323.684-322.309-319.041-310.285-295.471-278.885-260.804-252.167
-244.008-238.369 -227.82-207.378 -178.04-177.293-150.336-120.908 -93.104 -67.393
  -41.93 -15.292 -15.292 -13.797 -13.797  12.851  12.851  14.345  14.345  33.183
  50.208  67.034   89.01 111.863 139.487 171.804 198.831 224.473 227.939 229.444
  230.36 236.068 236.357 236.536 236.676 240.163 245.064 245.821 247.843 249.696
 253.263 254.827 255.942 257.108 259.628 260.057 261.202 261.312
  965.61  965.48   965.2  965.17  964.82  964.33  964.31  964.15  963.82  962.67
  962.55   962.5  961.81  960.86  960.06  959.79  959.77  959.54  958.76  958.49
  957.97  957.72  957.32  955.72   955.6  955.58  955.56  955.24  955.18  955.13
  954.63  954.57  954.55  954.49  954.32  953.81  953.09  952.66  952.26  952.08
  951.99  951.92  951.78   951.7  951.37  951.36  951.11  950.86  950.72  950.97
  951.58  951.75  952.75  952.75  952.75  952.99  952.99  952.99  952.01  952.54
  952.81     953  953.38  954.12  954.95   956.6  958.81  962.92  963.24  963.65
  963.86  964.99  965.04  965.09  965.11   965.8  966.85     967   967.4  967.76
  968.26  968.46  968.49  968.53  968.52  968.56  968.53  968.52
                                                                                
                                                                                
                                                                                
                                                                                
                                                                                
                                  950.12  950.48
                                                                                
                                                                                
                                                                
BR Coef=-1 , 1 , 0 ,, 0 ,,,0.8,0,1.2,0,
WSPro=,,,, 1 ,,,, 0 ,,,, 0 ,,,,-1 ,-1 ,-1 , 0 , 0 , 0 , 0 , 0
BC Design=,, 0 ,, 0 ,,,,,,
BC Use User HTab Curves=0
BC User HTab FreeFlow(D)= 0

Type RM Length L Ch R = 1 ,52495.01,266.9324,292.8095,286.3088
BEGIN DESCRIPTION:
SE. of Midway RD (TWE_28) - DS
END DESCRIPTION:
XS GIS Cut Line= 4
   1489706.00197    1131430.4439   1489576.04495    1131552.7021
    1489423.7769   1131709.37828   1489238.64304   1131895.33465
#Sta/Elev= 30
 -395.19  967.67-377.388  963.99-363.312  960.26-340.171  955.68-305.115  952.89
-255.903  951.56 -82.435  949.41 -43.414  949.82  -36.62  950.36  -26.21  949.84
 -23.311  948.79 -14.714  947.98 -11.665  947.31  -8.019  946.49  -4.573   944.5
   -.269  943.96   3.447  946.11   8.567  947.22  12.602  947.43  21.568  951.23
  31.799  951.29 115.887  953.27 177.363  956.44 191.558  957.56 209.051  960.25
 224.871  961.58 239.276  965.16 246.439  967.95 251.798  968.02 261.601  968.55
#Mann= 7 ,-1,0
 -395.19     .13       0-255.903      .1       0 -14.714     .12       0
 -11.665    .045       0  12.602     .12       0  31.799      .1       0
 251.798     .06       0
#XS Ineff= 2 , 0
       0     -30     952      30       0     952
Permanent Ineff=
       F       F
Bank Sta=-11.665,12.602
XS Rating Curve= 0 ,0
Skew Angle= 5
Exp/Cntr=0.5,0.3

Type RM Length L Ch R = 1 ,52202.20,580.3328,604.5864,567.6392
XS GIS Cut Line= 3
   1489569.14961    1131224.1063   1489243.62795   1131491.03412
   1488978.87073    1131710.2185
#Sta/Elev= 30
 -415.99  983.24 -398.56  978.25 -371.41  968.41  -336.7  957.25 -321.33  951.15
 -307.61  949.14 -162.64  948.88 -146.12  949.58 -134.36     949 -124.73  949.66
   -90.5  949.64  -34.79  948.91  -19.38  950.22  -11.56  948.54   -7.27  944.97
   -4.59  943.53    -.27  942.99    3.46  945.14    7.89  946.15   19.92  947.77
   29.17  950.83   45.66  951.02   156.3  954.36  237.03  958.43  241.47  959.11
  253.75  964.03  268.93  964.66   287.7  963.93  316.36  965.58  348.69  969.64
#Mann= 6 ,-1,0
 -415.99    .135       0   -7.27    .045       0    7.89     .13       0
   45.66      .1       0  253.75     .06       0   287.7     .14       0
Bank Sta=-7.27,7.89
XS Rating Curve= 0 ,0
Exp/Cntr=0.3,0.1

Type RM Length L Ch R = 1 ,51597.62,477.8195,544.9846,510.2537
XS GIS Cut Line= 3
   1489122.10039   1130826.97014   1488825.57119   1131107.73031
   1488659.85958   1131267.50919
#Sta/Elev= 30
 -408.59  978.15 -383.11     979 -361.59  975.05 -334.64  965.25 -312.43  954.81
 -295.09  948.17 -128.75  946.75  -33.94  948.63  -26.98  947.74  -19.68  945.51
   -12.9  945.27  -11.49   943.4   -6.33     941    4.04  941.92    5.72  943.36
    7.54  944.88   18.11  948.65   56.01  949.64      87  952.23   98.42  955.42
   117.8  956.25  124.21  958.31   130.8  962.33  157.96  968.61  183.86  968.35
   203.1   966.4  208.26  966.85  216.66  972.84  226.37  980.17  229.96  980.59
#Mann= 5 ,-1,0
 -408.59    .135       0  -11.49     .04       0    5.72      .1       0
  183.86     .06       0  216.66     .14       0
Bank Sta=-11.49,5.72
XS Rating Curve= 0 ,0
Exp/Cntr=0.3,0.1

Type RM Length L Ch R = 1 ,51052.63,267.2786,370.5237,365.7625
XS GIS Cut Line= 3
    1488853.0023   1130477.57677   1488484.07808   1130735.82415
   1488316.97703   1130859.52231
#Sta/Elev= 30
 -454.55   970.4  -401.9  959.34 -377.18  955.67 -352.64  953.24 -340.88  948.66
 -338.07  949.15 -320.45   947.2 -289.82  946.19 -279.69  946.95 -211.96945.2222
 -176.86  946.39 -143.77  945.72  -18.37  946.74   -9.99  945.15   -7.49   942.4
   -2.33     940    8.04  940.929.719999  942.36   11.54  943.88   20.15  946.96
      65  947.73   97.07950.1932  101.64  951.46  110.64  955.91  129.46  957.52
   138.7  961.42     146  963.34  158.57   964.2  193.76   969.3  203.69  969.78
#Mann= 5 ,-1,0
 -454.55    .135       0 -211.96     .13       0   -7.49     .04       0
9.719999     .13       0   97.07     .13       0
#XS Ineff= 1 ,-1
 -382.35 -298.78  952.67
Permanent Ineff=
       F
Bank Sta=-7.49,9.719999
XS Rating Curve= 0 ,0
Exp/Cntr=0.3,0.1

Type RM Length L Ch R = 1 ,50682.11,326.1364,434.0806,224.7923
BEGIN DESCRIPTION:
TWE_27X
END DESCRIPTION:
XS GIS Cut Line= 3
   1488695.59252   1130367.49869   1488395.77428    1130407.1332
   1488208.02362   1130428.22802
#Sta/Elev= 30
 -302.81   968.6 -270.56  963.23 -255.47  958.88 -224.94  954.75 -216.81  951.15
 -207.62   949.4 -196.52  950.76 -179.41  948.26 -137.45   945.2    -125  945.18
  -61.69  944.86  -42.05   942.6  -32.04  944.67  -22.21  945.09  -13.84  943.22
  -11.49  941.47   -6.33  939.07    4.04  939.99    5.72  941.43   11.81  944.85
   17.33  946.12   47.41   945.4   78.71   946.1   94.08  947.23  105.84  951.84
  110.16  954.06  128.65  955.11  137.51  959.94  159.47  966.26  188.55  971.53
#Mann= 5 ,-1,0
 -302.81    .135       0    -125     .13       0  -11.49     .04       0
    5.72     .13       0  105.84     .13       0
#XS Ineff= 2 , 0
         -198.26  951.57
Permanent Ineff=
       F       F
Bank Sta=-11.49,5.72
XS Rating Curve= 0 ,0
Exp/Cntr=0.3,0.1

Type RM Length L Ch R = 1 ,49759.58,514.6816,574.8795,496.1618
XS GIS Cut Line= 3
   1488239.93701   1129537.90518   1488001.17782   1129804.57218
   1487777.69619   1130054.39895
#Sta/Elev= 30
 -356.99  985.24 -345.69  981.09 -326.82  971.56 -289.38  951.88 -281.36  945.83
 -274.06  945.88 -260.83  943.69    -246  943.41 -207.57  943.93 -155.19  942.85
  -85.92  944.43  -44.97  942.97  -23.02  943.71  -20.88  943.36  -13.68  939.14
  -11.49  938.86   -6.33  936.46    4.04  937.38    5.72  938.82   18.66  944.12
   37.86943.6053   62.69  943.66   91.78  945.44  176.34  946.19  219.15  947.92
  255.02  950.62  284.33955.4391  293.79  956.05  306.26  960.15  336.14  966.58
#Mann= 5 ,-1,0
 -356.99     .14       0  -11.49     .04       0    5.72     .14       0
   37.86      .1       0  284.33     .14       0
#XS Ineff= 1 ,-1
 -327.79 -225.56  950.71
Permanent Ineff=
       F
Bank Sta=-11.49,5.72
XS Rating Curve= 0 ,0
Exp/Cntr=0.3,0.1

Type RM Length L Ch R = 1 ,48667.24,459.8952,475.5148,473.1491
XS GIS Cut Line= 3
   1487250.35171   1129112.55676   1487186.11549   1129208.91142
   1487001.21916   1129491.02986
#Sta/Elev= 30
 -117.05  960.72  -95.89  957.46  -79.01  955.58  -71.67  952.85  -62.76  950.58
  -46.17  943.06  -38.27  942.02  -19.33   941.5  -15.22  940.66  -14.77  936.09
    -3.6  933.96    6.06  933.17   14.34  934.49   15.44  936.02   19.18  941.09
   23.31  941.29   42.11  939.08   49.62  938.97   68.49  940.63  162.84  941.09
  201.79   942.2  234.63  944.51  246.91   946.8  267.31  948.45  280.41  954.68
  283.83  955.71  296.06  958.24  304.22  961.14  320.86  964.17  336.06  967.66
#Mann= 5 ,-1,0
 -117.05     .14       0  -14.77     .04       0   15.44     .14       0
   68.49      .1       0  246.91     .14       0
Bank Sta=-14.77,15.44
XS Rating Curve= 0 ,0
Exp/Cntr=0.3,0.1

Type RM Length L Ch R = 1 ,47777.40,468.511,425.6777,370.561
XS GIS Cut Line= 3
   1486764.02231   1128491.89567   1486609.07415   1128629.91699
   1486334.33432   1128842.15682
#Sta/Elev= 30
  -212.4   955.9 -148.15   951.6 -112.73  947.96   -92.3  946.59  -54.59  942.05
  -21.47  941.31  -18.25  940.93  -17.65  938.02  -15.86     936  -14.55  934.41
    -3.6  932.54    6.06  931.75   14.34  933.07   16.57  935.98   16.57  936.03
   19.22  939.63   42.34  938.07  115.31  938.96  174.93  941.36  193.82  942.41
  201.21  943.96  211.64  947.43  224.87  948.16   233.1  951.42  266.31  956.36
  274.13  958.61   300.4  960.26   318.9   962.6  331.74  965.33  342.28  965.68
#Mann= 6 ,-1,0
  -212.4     .14       0  -15.86     .04       0   16.57     .14       0
   42.34      .1       0  174.93     .14       0  266.31      .1       0
Bank Sta=-15.86,16.57
XS Rating Curve= 0 ,0
Exp/Cntr=0.3,0.1

Type RM Length L Ch R = 1 ,47351.72,223.5139,243.5831,252.1278
BEGIN DESCRIPTION:
TWE_26X
END DESCRIPTION:
XS GIS Cut Line= 4
   1486278.34449   1128257.52034   1486278.29724   1128391.04462
   1486275.74016     1128478.875   1486118.18766   1128528.35433
#Sta/Elev= 30
 -132.37  982.22 -119.24  978.42 -103.55  972.08  -81.43  964.76  -65.51  952.44
  -49.39  952.37  -45.33  951.45  -44.01  950.76   -43.9  949.98  -27.24  941.63
   -19.2  938.58  -14.77  933.59    -3.6  931.46    6.06  930.67   13.93  931.89
   20.38  935.81   29.03  938.07   36.87  938.13   79.22   940.9   79.64  941.45
   85.77   941.1   89.02  939.98   93.93  941.34   98.42  941.78  111.37   941.8
  132.57  946.06  147.72  946.62  156.08  950.31  228.95     959  254.16  963.86
#Mann= 3 ,-1,0
 -132.37     .13       0  -14.77     .04       0   13.93     .13       0
#XS Ineff= 2 , 0
                           80.12          950.95
Permanent Ineff=
       F       F
Bank Sta=-14.77,13.93
XS Rating Curve= 0 ,0
Exp/Cntr=0.3,0.1

Type RM Length L Ch R = 1 ,46320.07,355.7927,668.618,610.6862
XS GIS Cut Line= 4
   1485380.84941   1127792.95899   1485379.57185   1127937.06726
   1485379.11319    1128128.0292   1485444.48228   1128207.20899
#Sta/Elev= 30
 -143.32  960.53 -120.76  959.25 -102.96  956.95  -73.09  949.74  -59.27  945.18
  -47.81  937.15  -39.37  937.55  -24.83   936.7  -18.44   933.9   -9.43  932.66
   -9.17  927.49   -4.18     928     .28  930.94     8.8  933.09   27.88  936.15
    39.2   936.1   53.54  934.97   60.45  934.96   82.32  937.39  106.58  938.92
  121.29  938.37  130.33  938.64  169.23  940.49  178.52  941.76  182.38  941.17
  189.58  941.47  201.39  944.16  232.91  949.13  274.41  953.74  294.43  956.64
#Mann= 3 ,-1,0
 -143.32     .13       0   -9.43     .04       0     8.8     .13       0
#XS Ineff= 2 , 0
                          107.42          948.64
Permanent Ineff=
       F       F
Bank Sta=-9.43,8.8
XS Rating Curve= 0 ,0
Exp/Cntr=0.3,0.1

Type RM Length L Ch R = 1 ,45651.45,594.5614,684.3304,641.0182
XS GIS Cut Line= 3
   1485248.56266    1127619.9101    1484906.6145   1128163.62927
   1484787.67585   1128847.52559
#Sta/Elev= 30
    -642  977.44 -549.45  972.73 -470.79  960.65 -419.48  955.09 -388.91  954.45
 -379.49  952.55 -365.67  947.16 -357.98  941.92 -333.47  941.96 -324.59   938.2
 -303.25  935.04 -234.06  935.26 -164.41  932.26     -76  933.71   -9.89  932.27
   -9.43   931.1   -9.17  926.43   11.24  932.12    19.5  933.13   59.16  931.94
  141.93   931.5  256.22   934.4  391.24   941.7  493.77  944.63  591.71  952.27
  660.24  953.19  666.64  954.99  681.75  962.92  686.42   964.3  694.47  963.51
#Mann= 4 ,-1,0
    -642     .14       0   -9.89    .045       0   11.24     .14       0
   59.16      .1       0
#XS Ineff= 2 , 0
       0                     170       0     945
Permanent Ineff=
       F       F
Bank Sta=-9.89,11.24
XS Rating Curve= 0 ,0
Exp/Cntr=0.5,0.3
